--- CDC_Consolidated_Model.prj (project) ---

Proj Title=Upper Trinity CDC Consolidated Model
Current Plan=p11
Default Exp/Contr=0.3,0.1
English Units
Geom File=g01
Geom File=g02
Geom File=g03
Geom File=g04
Geom File=g11
Geom File=g12
Geom File=g13
Flow File=f01
Flow File=f02
Flow File=f03
Flow File=f04
Flow File=f05
Flow File=f06
Flow File=f11
Flow File=f12
Flow File=f13
Plan File=p01
Plan File=p02
Plan File=p03
Plan File=p04
Plan File=p05
Plan File=p06
Plan File=p11
Plan File=p12
Plan File=p13
Y Axis Title=Elevation
X Axis Title(PF)=Main Channel Distance
X Axis Title(XS)=Station
BEGIN DESCRIPTION:
Upper Trinity River CDC Consolidated Model
For each new update of the CDC Consolidated Model, enter date here: 1 December 2025
Previous versions: 24 September 2024
                                12 August 2024
                                  22 July 2024
                                  19 July 2024
                                 1 March 2024
                               16 February 2024
                               30 October 2023
                               24 October 2023
                                01 August 2023
                             14 February 2023
Note:  Run the NFIP-CDC Model using HEC-RAS version 6.1 or newer.
--------------------------------------------------------------------------------------------------------------------------------------------
Developed by the Federal Emergency Management Agency (FEMA) Region 6 and the US Army Corps of Engineers - Fort Worth District (USACE).  The Upper Trinity River CDC Consolidated Model represents the upper Trinity River FEMA Existing Model (plans 01 - 06) and the upper Trinity River CDC Model (plans 11 - 13) under one project (.prj) file.
The model was shared with the NCTCOG Trinity Flood Management Task Force (FMTF) for review in February 2023.  Iinformation regarding the Upper Trinity River CDC Consolidated Model Model and the CDC program can be found at the following website: http://trinityrivercdc.com/
--------------------------------------------------------------------------------------------------------------------------------------------
CDC Model Disclaimer: The Corridor Development Certificate (CDC) Model, updated as of 14 February 2023.  The model includes CDC granted projects as of January 2022 (both constructed and not constructed).  The model includes future conditions (2055) upper Trinity River watershed flows.  Projects that been granted a CDC since 2022 will be incorporated in future model updates.
Existing Model Disclaimer: This is a FEMA preliminary model, updated as of 14 February 2023.  This model is not yet a regulatory/effective model and is subject to change without notice.  The end user bears the responsibility for ensuring use of the most appropriate and current model. The NFIP effective model with tie-ins will need to be submitted in conjunction with this updated model.  Includes constructed CDC project geometries that have gone through the FEMA Letter of Map Change (LOMC) process.  Note that FEMA will require the submittal of the effective model (with appropriate tie-ins) in addition to the preliminary model for any formal map change requests - until the preliminary model becomes effective.  The NFIP Model includes existing conditions upper Trinity River watershed flows.
--------------------------------------------------------------------------------------------------------------------------------------------
AEP (Annual Exceedance Probability) equivalencies:
0.2%  500-year flood
1%     100-year flood
2%       50-year flood
4%       25-year flood
10%     10-year flood
20%       5-year flood
50%       2-year flood
River designations:
CF         Clear Fork Trinity River
EF            Elm Fork Trinity River
WF        West Fork Trinity River
TRMS    Trinity River main stem
END DESCRIPTION:
DSS Export Rating Curves= 0
DSS Export Rating Curve Sorted= 0
DSS Export Volume Flow Curves= 5
Main Stem       ,ms              ,148136. ,ms              ,120629.
Main Stem       ,ms              ,120629. ,ms              ,108276
Main Stem       ,ms              ,108276  ,ms              ,82361
Main Stem       ,ms              ,82361   ,ms              ,75882
Main Stem       ,ms              ,75882   ,ms              ,51060
DXF Filename=..\..\..\..\..\..\TempKdrive\Danella\Work\CDC\CDC Model\CDC-2012 working\working- use this!\2012 november 29 submitted to nctcog\UTCDC-1-2012.
DXF OffsetX= 0
DXF OffsetY= 0
DXF ScaleX= 1
DXF ScaleY= 10
Specific Locations Profile Table=SplitFlow_2to100                     , 15
Elm Fork        ,ef5             ,139643
Elm Fork        ,ef4             ,138514
Elm Fork Split2 ,efs2            ,132950
Elm Fork        ,ef3             ,49916
Elm Fork        ,ef2             ,48911
Elm Fork Split1 ,efs1            ,9111
West Fork       ,wf3             ,112574
West Fork       ,wf3f            ,111680
West Fork       ,wf3e            ,111679
West Fork       ,wf3d            ,85875
West Fork       ,wf3b            ,84548
West Fork       ,wf3c            ,84549
West Fork       ,wf3a            ,55761
West Fork       ,wf2             ,53730
West Fork Split ,wfs             ,54405
Specific Locations Profile Table=SplitFlow_500_SPF                    , 3
Elm Fork        ,PGBT split west ,97178
Elm Fork        ,PGBT split east ,97178.1
Elm Fork        ,ef3             ,97919
Specific Locations Profile Table=SplitFlow_500toSPF                   , 6
Elm Fork        ,PGBT split west ,97178
Elm Fork        ,PGBT split east ,97178.1
Elm Fork        ,ef3             ,97919
Elm Fork        ,ef5             ,139643
Elm Fork        ,ef4             ,138514
Elm Fork Split2 ,efs2            ,132950
Specific Locations Profile Table=EF3-81856                            , 4
Elm Fork        ,ef3             ,82779
Elm Fork        ,ef3             ,81865
Elm Fork        ,ef3             ,80596
Elm Fork        ,ef3             ,78205
Specific Locations Profile Table=ef3_FW                               , 11
Elm Fork        ,ef3             ,97191
Elm Fork        ,ef3             ,93954
Elm Fork        ,ef3             ,93374
Elm Fork        ,ef3             ,93324
Elm Fork        ,ef3             ,93273
Elm Fork        ,ef3             ,93211
Elm Fork        ,ef3             ,93208
Elm Fork        ,ef3             ,93207
Elm Fork        ,ef3             ,93206
Elm Fork        ,ef3             ,93205
Elm Fork        ,ef3             ,93155

--- CDC_Consolidated_Model.p11 (plan) ---

Plan Title=CDC: 50% to 0.2% AEP, SPF [WF/CF]
Program Version=5.07
Short Identifier=CDC Plan 11
Geom File=g11
Flow File=f11
Subcritical Flow
K Sum by GR= 0
Std Step Tol= 0.01
Critical Tol= 0.01
Num of Std Step Trials= 20
Max Error Tol= 0.3
Flow Tol Ratio= 0.001
Split Flow NTrial= 30
Split Flow Tol= 0.02
Split Flow Ratio= 0.02
Log Output Level= 0
Friction Slope Method= 1
Unsteady Friction Slope Method= 2
Unsteady Bridges Friction Slope Method= 1
Parabolic Critical Depth
Global Vel Dist= 0 , 0 , 0
Global Log Level= 0
CheckData=True
Encroach Param=-1 ,0,0, 0
BEGIN DESCRIPTION:
CDC Model
This plan is valid upstream of West Fork cross-section 206218 for the West Fork and Clear Fork.  This plan represents the 50%, 20%, 10%, 4%, 2%, 1%, 0.2% AEP and SPF peak flows and geometry.
END DESCRIPTION:
Computation Interval=1HOUR
Output Interval=1HOUR
Instantaneous Interval=1HOUR
Mapping Interval=1HOUR
Computation Time Step Use Courant=        0
Computation Time Step Use Time Series=    0
Computation Time Step Count To Double=0
Computation Time Step Max Doubling=0
Computation Time Step Max Halving=0
Computation Time Step Residence Courant=0
Run HTab= 0
Run UNet= 0
Run Sediment= 0
Run PostProcess= 0
Run WQNet= 0
Run RASMapper= 0
UNET Theta= 1
UNET Theta Warmup= 1
UNET ZTol= 0.02
UNET ZSATol= 0.05
UNET MxIter= 20
UNET Max Iter WO Improvement= 0
UNET MaxInSteps= 0
UNET DtIC= 0
UNET DtMin= 0
UNET MaxCRTS= 20
UNET WFStab= 2
UNET SFStab= 1
UNET WFX= 1
UNET SFX= 1
UNET 1D Methodology=Finite Difference
UNET DSS MLevel= 4
UNET Pardiso=0
UNET DZMax Abort= 100
UNET Use Existing IB Tables=-1
UNET Froude Reduction=False
UNET Froude Limit= 1
UNET Froude Power= 10
UNET D1 Cores= 0
UNET D2 Coriolis=0
UNET D2 Cores= 0
UNET D2 Theta= 1
UNET D2 Theta Warmup= 1
UNET D2 Z Tol= 0.01
UNET D2 Volume Tol= 0.01
UNET D2 Max Iterations= 20
UNET D2 Equation= 0
UNET D2 RampUpFraction=0.1
UNET D2 TimeSlices= 1
UNET D2 BCVolumeCheck=0
UNET D1D2 MaxIter= 0
UNET D1D2 ZTol=0.01
UNET D1D2 QTol=0.1
UNET D1D2 MinQTol=1
Write IC File= 0
Write IC File at Fixed DateTime=0
Write IC File at Sim End=0
Echo Input=False
Echo Parameters=False
Echo Output=False
Write Detailed= 0
HDF Write Warmup=0
HDF Write Time Slices=0
HDF Flush=0
HDF Face Node Velocities=0
HDF Compression= 1
HDF Chunk Size= 1
HDF Spatial Parts= 1
HDF Use Max Rows=0
HDF Fixed Rows= 1
Calibration Method= 0
Calibration Iterations= 20
Calibration Max Change=0.05
Calibration Tolerance=0.2
Calibration Maximum=1.5
Calibration Minimum=0.5
Calibration Optimization Method= 1
WQ AD Non Conservative
WQ ULTIMATE=-1
WQ Max Comp Step=1HOUR
WQ Output Interval=15MIN
WQ Output Selected Increments= 0
WQ Output face flow=0
WQ Output face velocity=0
WQ Output face area=0
WQ Output face dispersion=0
WQ Output cell volume=0
WQ Output cell surface area=0
WQ Output cell continuity=0
WQ Output cumulative cell continuity=0
WQ Output face conc=0
WQ Output face dconc_dx=0
WQ Output face courant=0
WQ Output face peclet=0
WQ Output face adv mass=0
WQ Output face disp mass=0
WQ Output cell mass=0
WQ Output cell source sink temp=0
WQ Output nsm pathways=0
WQ Output nsm derived pathways=0
WQ Output MaxMinRange=-1
WQ Daily Max Min Mean=-1
WQ Daily Range=0
WQ Daily Time=0
WQ Create Restart=0
WQ Fixed Restart=0
WQ System Summary=0
WQ Write To DSS=0
WQ Use Fixed Temperature=0
Sorting and Armoring Iterations= 10
XS Update Threshold= 0.02
Bed Roughness Predictor= 0
Hydraulics Update Threshold= 0.02
Energy Slope Method= 0
Volume Change Method= 0
Sediment Retention Method= 0
XS Weighting Method= 0
Number of US Weighted Cross Sections= 1
Number of DS Weighted Cross Sections= 1
Upstream XS Weight=0.25
Main XS Weight=0.5
Downstream XS Weight=0.25
Number of DS XS's Weighted with US Boundary= 1
Upstream Boundary Weight= 1
Weight of XSs Associated with US Boundary= 0
Number of US XS's Weighted with DS Boundary= 1
Downstream Boundary Weight= 0.5
Weight of XSs Associated with DS Boundary= 0.5
Percentile Method= 0
Sediment Output Level= 4
Mass or Volume Output= 0
Output Increment Type= 1
Profile and TS Output Increment= 10
XS Output Flag= 0
XS Output Increment= 10
Write Gradation File= 0
Read Gradation Hotstart= 0
Write HDF5 File= 1
Write Binary Output= 1
Write DSS Sediment File= 0
SV Curve= 0
Specific Gage Flag= 0

--- CDC_Consolidated_Model.p01 (plan) ---

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Plan Title=Exist: 10%, 4%, 2%, 1% AEP [WF/EF/TRMS]
Program Version=6.60
Short Identifier=Existing Plan 1
Geom File=g01
Flow File=f01
Secant Critical Depth
Flow Ratio Tolerance=0.1
Flow Ratio Min Ratio=0.5
Flow Ratio Max Ratio=4
Flow Ratio Max Iterations= 10
Existing Model
This plan is valid downstream of West Fork cross-section 206218 for the West Fork, Elm Fork, and Trinity River Main Stem.  This plan represents the 10%, 4%, 2%, 1% AEP peak flows and geometry.
UNET Gravity=32.17405
UNET WindReference=Eulerian
UNET WindDragFormulation=Hsu (1988)
UNET D2 Advanced Convergence=0
UNET D2 WS Max Tol=0.15
UNET D2 WS RMS Tol=0.002
UNET D2 WS Stall Tol=1
UNET D2 Turbulence Formulation=Non-Conservative (original)
UNET D2 Eddy Viscosity=0.3
UNET D2 Transverse Eddy Viscosity=0.3
UNET D2 Smagorinsky Mixing=0
UNET D2 Cores=0
UNET D2 SolverType=PARDISO (Direct)
UNET D2 Minimum Iterations= 3
UNET D2 Maximum Iterations= 30
UNET D2 Restart Number= 10
UNET D2 Relaxation Coeff=1.3
UNET D2 SOR Precondition Iterations= 10
UNET D2 ILUT Maximum Fill= 8
UNET D2 ILUT Tolerance=1E-08
UNET D2 Convergence Tolerance=0.00001
PS Theta= 1
PS WS Tol= 0.01
PS Volume Tol= 0.01
PS Max Iterations= 20
PS Equation= 0
PS Advance Time Step=-1
PS Target Courant=0.9
PS Time Slices= 1
PS Iterate With 2D=0
PS Project Initial WSE from DS=-1
PS Ramp Up Initial WSE from US=-1
PS Cores=0
DSS File=dss
Processes Affected by Predictor=Sediment Only
Energy Slope Method= 2
Sediment TS Multiplier= 1
Warm Up Method= 0
Transport Output Increment 1
Read HDF5 Sediment Hotstart= 0
Sediment Hotstart Type= 0
DSS Sediment Output Type= 1
Subcell Erosion Methods= 0
Subcell Deposition Methods= 0
Advection Scheme= 1
Matrix Solver= 0
Implicit Weighting Factor= 1
Maximum Outer Loop Convergence Iterations= 5
Convergence Maximum Absolute= 0.001
Convergence RMSE= 0.0001
Grain Fractions Max Abs Error= 0.001
Max Subgrid Regions= 1
Max Subgrid Length Scale= 3.402823E+38
Initial Layer Thickness= 3
Min Layer Thickness= 0.1
Max Layer Thickness= 6
Number of Layers= 5

--- CDC_Consolidated_Model.p02 (plan) ---

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Plan Title=Exist: 0.2% AEP [WF/EF/TRMS]
Program Version=6.60
Short Identifier=Existing Plan 2
Geom File=g02
Flow File=f02
Flow Ratio Tolerance=0.1
Flow Ratio Min Ratio=0.5
Flow Ratio Max Ratio=4
Flow Ratio Max Iterations= 10
Existing Model
This plan is valid downstream of West Fork cross-section 206218 for the West Fork, Elm Fork, and Trinity River Main Stem.  This plan represents the 0.2% AEP peak flows and geometry.
UNET Gravity=32.17405
UNET WindReference=Eulerian
UNET WindDragFormulation=Hsu (1988)
UNET D2 Advanced Convergence=0
UNET D2 WS Max Tol=0.15
UNET D2 WS RMS Tol=0.002
UNET D2 WS Stall Tol=1
UNET D2 Turbulence Formulation=Non-Conservative (original)
UNET D2 Eddy Viscosity=0.3
UNET D2 Transverse Eddy Viscosity=0.3
UNET D2 Smagorinsky Mixing=0
UNET D2 Cores=0
UNET D2 SolverType=PARDISO (Direct)
UNET D2 Minimum Iterations= 3
UNET D2 Maximum Iterations= 30
UNET D2 Restart Number= 10
UNET D2 Relaxation Coeff=1.3
UNET D2 SOR Precondition Iterations= 10
UNET D2 ILUT Maximum Fill= 8
UNET D2 ILUT Tolerance=1E-08
UNET D2 Convergence Tolerance=0.00001
PS Theta= 1
PS WS Tol= 0.01
PS Volume Tol= 0.01
PS Max Iterations= 20
PS Equation= 0
PS Advance Time Step=-1
PS Target Courant=0.9
PS Time Slices= 1
PS Iterate With 2D=0
PS Project Initial WSE from DS=-1
PS Ramp Up Initial WSE from US=-1
PS Cores=0
DSS File=dss
Processes Affected by Predictor=Sediment Only
Energy Slope Method= 2
Sediment TS Multiplier= 1
Warm Up Method= 0
Transport Output Increment 1
Read HDF5 Sediment Hotstart= 0
Sediment Hotstart Type= 0
DSS Sediment Output Type= 1
Subcell Erosion Methods= 0
Subcell Deposition Methods= 0
Advection Scheme= 1
Matrix Solver= 0
Implicit Weighting Factor= 1
Maximum Outer Loop Convergence Iterations= 5
Convergence Maximum Absolute= 0.001
Convergence RMSE= 0.0001
Grain Fractions Max Abs Error= 0.001
Max Subgrid Regions= 1
Max Subgrid Length Scale= 3.402823E+38
Initial Layer Thickness= 3
Min Layer Thickness= 0.1
Max Layer Thickness= 6
Number of Layers= 5

--- CDC_Consolidated_Model.p03 (plan) ---

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Plan Title=Exist: 10%,4%,2%,1%,0.2%,1%+ AEP [WF/CF]
Program Version=6.60
Short Identifier=Existing Plan 3
Geom File=g03
Flow File=f03
Flow Ratio Tolerance=0.1
Flow Ratio Min Ratio=0.5
Flow Ratio Max Ratio=4
Flow Ratio Max Iterations= 10
Existing Model
This plan is valid upstream of West Fork cross-section 206218 for the West Fork and Clear Fork.  This plan represents the 10%, 4%, 2%, 1%, 0.2%, 1%+ AEP peak flows and geometry.
UNET Gravity=32.17405
UNET WindReference=Eulerian
UNET WindDragFormulation=Hsu (1988)
UNET D2 Advanced Convergence=0
UNET D2 WS Max Tol=0.15
UNET D2 WS RMS Tol=0.002
UNET D2 WS Stall Tol=1
UNET D2 Turbulence Formulation=Non-Conservative (original)
UNET D2 Eddy Viscosity=0.3
UNET D2 Transverse Eddy Viscosity=0.3
UNET D2 Smagorinsky Mixing=0
UNET D2 Cores=0
UNET D2 SolverType=PARDISO (Direct)
UNET D2 Minimum Iterations= 3
UNET D2 Maximum Iterations= 30
UNET D2 Restart Number= 10
UNET D2 Relaxation Coeff=1.3
UNET D2 SOR Precondition Iterations= 10
UNET D2 ILUT Maximum Fill= 8
UNET D2 ILUT Tolerance=1E-08
UNET D2 Convergence Tolerance=0.00001
PS Theta= 1
PS WS Tol= 0.01
PS Volume Tol= 0.01
PS Max Iterations= 20
PS Equation= 0
PS Advance Time Step=-1
PS Target Courant=0.9
PS Time Slices= 1
PS Iterate With 2D=0
PS Project Initial WSE from DS=-1
PS Ramp Up Initial WSE from US=-1
PS Cores=0
Processes Affected by Predictor=Sediment Only
Energy Slope Method= 2
Sediment TS Multiplier= 1
Warm Up Method= 0
Transport Output Increment 1
Read HDF5 Sediment Hotstart= 0
Sediment Hotstart Type= 0
DSS Sediment Output Type= 1
Subcell Erosion Methods= 0
Subcell Deposition Methods= 0
Advection Scheme= 1
Matrix Solver= 0
Implicit Weighting Factor= 1
Maximum Outer Loop Convergence Iterations= 5
Convergence Maximum Absolute= 0.001
Convergence RMSE= 0.0001
Grain Fractions Max Abs Error= 0.001
Max Subgrid Regions= 1
Max Subgrid Length Scale= 3.402823E+38
Initial Layer Thickness= 3
Min Layer Thickness= 0.1
Max Layer Thickness= 6
Number of Layers= 5
