HEC-RAS study CDC_Consolidated_Model.prj: Upper Trinity CDC Consolidated Model

--- CDC_Consolidated_Model.p04 (plan) ---

Plan Title=Exist: FEMA Floodway [WF/EF/TRMS]
Program Version=6.60
Short Identifier=Existing Plan 4
Geom File=g01
Flow File=f04
Subcritical Flow
K Sum by GR= 0
Std Step Tol= 0.01
Critical Tol= 0.01
Num of Std Step Trials= 20
Max Error Tol= 0.3
Flow Tol Ratio= 0.001
Split Flow NTrial= 30
Split Flow Tol= 0.02
Split Flow Ratio= 0.02
Log Output Level= 0
Friction Slope Method= 1
Unsteady Friction Slope Method= 2
Unsteady Bridges Friction Slope Method= 1
Parabolic Critical Depth
Global Vel Dist= 0 , 0 , 0
Global Log Level= 0
CheckData=True
Encroach Param=-1 ,0,0, 2
Encroach River=Elm Fork
Encroach Reach=ef6
Encroach Node=153340
       1    9797   10128
Encroach Node=153231
       1    9848    9999
Encroach Node=153202
       1    9863    9999
Encroach Node=153201
       1    9855    9991
Encroach Node=153103
       1    9823   10052
Encroach Node=152112
       1    3163    3423
Encroach Node=151332
       1    4440    4667
Encroach Node=150604
       1    5747    6064
Encroach Node=149605
       1    7273    7532
Encroach Node=148735
       1    8445    8674
Encroach Node=148113
       1    8212    8481
Encroach Reach=ef5
Encroach Node=147501
       1    6110    9580
Encroach Node=147401
       1    6140   10404
Encroach Node=147312
       1    6179   10454
Encroach Node=147311
       1    6190   10464
Encroach Node=147216
       1    6255   10517
Encroach Node=146384
       1    8750   12912
Encroach Node=146243
       1    3300    7444
Encroach Node=145841
       1    3400    7529
Encroach Node=145408
       1    3465    7799
Encroach Node=145103
       1    3664    8015
Encroach Node=144866
       1    3826    8090
Encroach Node=144665
       1    3566    7597
Encroach Node=144557
       1    2950    6840
Encroach Node=144486
       1   10336   14133
Encroach Node=144323
       1   10569   14108
Encroach Node=144156*
       1   10513   13916
Encroach Node=143767
       1   10274   13761
Encroach Node=143249*
       110435.65   13134
Encroach Node=142911
       1    9721   12554
Encroach Node=142659*
       1 9352.44   12229
Encroach Node=141707
       1    8105    9971
Encroach Node=141529
       1    7538    9245
Encroach Node=141407*
       1 7373.28    9062
Encroach Node=141309
       1 7245.05    8939
Encroach Node=139760
       1    6476    9270
Encroach Node=139655
       1    6303    9044
Encroach Reach=ef4
Encroach Node=138526
       1  7212.6  7438.6
Encroach Node=137889
       1  7507.5    7665
Encroach Node=137364
       1    7424    7583
Encroach Node=136161
       1    6336    6481
Encroach Node=135383
       1    5809    5964
Encroach Node=134552
       1    5458    5626
Encroach Node=133647
       1    4731    4979
Encroach Node=132670
       1    1854    2590
Encroach Node=132012
       1    1040    1344
Encroach Node=131546
       1    1860    2093
Encroach Node=130990
       1    1067    1791
Encroach Node=130391
       1    1298    1680
Encroach Node=129702
       1    1317    1677
Encroach Node=129061
       1    1280    1661
Encroach Node=128272
       1    1759    1973
Encroach Node=127699
       1    1297    1732
Encroach Node=127387
       1    1280    1633
Encroach Node=126832
       1    1348    1544
Encroach Node=126831
       1    1348    1544
Encroach Node=126288
       1    1130    1675
Encroach Node=126287
       1    1130    1675
Encroach Node=126185
       1    1040    1676
Encroach Node=126184
       1    1040    1676
Encroach Reach=ef3
Encroach Node=125671
       1    1045    2536
Encroach Node=124988
       1    1046    2650
Encroach Node=123537
       1    1020    3430
Encroach Node=123190
       1    1003    4340
Encroach Node=122933
       1     990    4740
Encroach Node=120765
       1     980    5515
Encroach Node=119726
       1    1071    6420
Encroach Node=118745
       1    4021   10560
Encroach Node=116394
       1    5000   11498
Encroach Node=113808
       1    7000   12500
Encroach Node=112738
       1    7377   12004
Encroach Node=112632
       1    7510   11872
Encroach Node=112622
       1    7510   11863
Encroach Node=112469
       1    7326   11790
Encroach Node=111948
       1    5740    9930
Encroach Node=110586
       1    2785    7156
Encroach Node=110488
       1    2600    7142
Encroach Node=110448
       1    2600    7142
Encroach Node=110398
       1    2620    7325
Encroach Node=110274
       1    2620    7325
Encroach Node=110227
       1    2609    7140
Encroach Node=110187
       1    2609    7140
Encroach Node=110088
       1    2600    6663
Encroach Node=109695
       1    1010    4691
Encroach Node=109459
       1    1070    4634
Encroach Node=109411
       1     260    3814
Encroach Node=109357
       1     255    3800
Encroach Node=107977
       1    1020    4419
Encroach Node=107870
       1     285    3719
Encroach Node=106693
       1    1025    5043
Encroach Node=106669
       1    1017    5074
Encroach Node=105948
       1    1823    6450
Encroach Node=105564*
       1    2090    6923
Encroach Node=105179
       1    2375    7265
Encroach Node=104984
       1    2151    7167
Encroach Node=104961*
       1    2123    7162
Encroach Node=102709
       1    1844    8255
Encroach Node=101441
       1    3008    8764
Encroach Node=99721
       1    3453    8400
Encroach Node=98898
       1    4030    8650
Encroach Node=97933
       1    4517    8600
Encroach Node=97191
       1    5351    8700
Encroach Node=93954
       1    7005    9220
Encroach Node=93374
       1    8000    9079
Encroach Node=93324
       1    8059    9090
Encroach Node=93211
       1    8059    9054
Encroach Node=93208
       1    8240    9075
Encroach Node=93207
       1    8277    9110
Encroach Node=93206
       1    8275    9104
Encroach Node=93205
       1    8275    9104
Encroach Node=93155
       1    8308    9102
Encroach Node=92366
       1    7664    8938
Encroach Node=91545
       1    7450    9706
Encroach Node=90547
       1    7530   10150
Encroach Node=89708
       1    7700   10332
Encroach Node=88727
       1    7800   11004
Encroach Node=88523
       1    6115   11436
Encroach Node=88009
       1    6177   11648
Encroach Node=87661
       1    6860   12215
Encroach Node=87553
       1    4930   10450
Encroach Node=87533
       1    4930   10450
Encroach Node=87532
       1    4930   10450
Encroach Node=87439
       1    4931   10184
Encroach Node=87354
       1    4931   10164
Encroach Node=87353
       1    4931   10164
Encroach Node=87207
       1    5010   10221
Encroach Node=86799
       1    4806    9970
Encroach Node=86633
       1    4535    9588
Encroach Node=86123
       1    4381    8750
Encroach Node=84978
       1    2530    6700
Encroach Node=84503
       1    1050    5130
Encroach Node=83547
       1    1098    5030
Encroach Node=82779
       1    1298    4950
Encroach Node=81865
       1    1274    4870
Encroach Node=80596
       1    1279    4790
Encroach Node=78205
       1    1050    4330
Encroach Node=76493
       1    1050    4310
Encroach Node=72731
       1    1077    4240
Encroach Node=71700
       1    1171    4170
Encroach Node=70611
       1    1148    4080
Encroach Node=69720
       1    1050    3850
Encroach Node=68724
       1    1300    3440
Encroach Node=67631
       1    1400    3170
Encroach Node=67494
       1    1550    3078
Encroach Node=67381
       1    1576    2937
Encroach Node=67283
       1    1576    2933
Encroach Node=67282
       1    1574    2932
Encroach Node=67188
       1    1539    2891
Encroach Node=66179
       1    1035    2874
Encroach Node=65332
       1    1015    2987
Encroach Node=64635
       1    1142    3094
Encroach Node=64504
       1    3761    5633
Encroach Node=64414
       1    3761    5633
Encroach Node=64413
       1    3761    5633
Encroach Node=64296
       1    3761    5633
Encroach Node=64211
       1    3761    5618
Encroach Node=64210
       1    3761    5617
Encroach Node=64124
       1    3678    5610
Encroach Node=63400
       1    3520    5925
Encroach Node=62370
       1    3246    5057
Encroach Node=61222
       1    3037    4031
Encroach Node=60829
       1    2833    3941
Encroach Node=59979
       1    2600    4078
Encroach Node=59087
       1    3214    4630
Encroach Node=58673
       1    3614    4751
Encroach Node=58631
       1    3651    4745
Encroach Node=58552
       1    3626    4722
Encroach Node=58448
       1    3564    4780
Encroach Node=58065
       1    3220    5000
Encroach Node=57214
       1    2400    5200
Encroach Node=55715
       1    1770    5303
Encroach Node=55003
       1    1372    5261
Encroach Node=54962
       1     992    4896
Encroach Node=54833
       1    1076    5024
Encroach Node=54781
       1    1104    5068
Encroach Node=54638
       1    1174    5199
Encroach Node=54493
       1    1263    5350
Encroach Node=54428
       1    1309    5422
Encroach Node=54251
       1    1249    5428
Encroach Node=53311
       1    1293    5570
Encroach Node=52413
       1    1351    5230
Encroach Node=51531
       1    1126    4650
Encroach Node=50772
       1    1320    4540
Encroach Node=49936
       1    1434    4550
Encroach Reach=ef2
Encroach Node=48931
       1    2202    4769
Encroach Node=48820
       1    2352    4839
Encroach Node=48731
       1    2320    4821
Encroach Node=48730
       1    2320    4823
Encroach Node=48630
       1    2290    4905
Encroach Node=47811
       1    2261    4989
Encroach Node=44365
       1    1403    3500
Encroach Node=44320
       1    1415    3210
Encroach Node=44319
       1    1414    3195
Encroach Node=44314
       1    1401    3168
Encroach Node=44313
       1    1411    3175
Encroach Node=44263
       1    1350    3145
Encroach Node=43164
       1    2085    4290
Encroach Node=43054
       1    2020    4400
Encroach Node=43008
       1    2002    4370
Encroach Node=42902
       1    1950    4310
Encroach Node=40798
       1    2350    4674
Encroach Node=39841
       1    2500    5312
Encroach Node=37472
       1    1769    4797
Encroach Node=37336
       1    1830    4803
Encroach Node=37317
       1    1837    4803
Encroach Node=37316
       1    1838    4803
Encroach Node=37191
       1    1845    4776
Encroach Node=36129
       1    2114    4600
Encroach Node=35426
       1    2084    4753
Encroach Node=34376
       1    2126    5238
Encroach Node=34342
       1    2139    5270
Encroach Node=34222
       1    2212    5349
Encroach Node=34197
       1    2224    5363
Encroach Node=34196
       1    2224    5363
Encroach Node=34101
       1    2274    5421
Encroach Node=34037
       1    2338    5455
Encroach Node=32771
       1    3290    6470
Encroach Node=31903
       1    3361    6673
Encroach Reach=ef1
Encroach Node=31628
       1    3349    6688
Encroach Node=30779
       1    3700    6489
Encroach Node=29562
       1    4400    6224
Encroach Node=29459
       1    4345    6180
Encroach Node=29341
       1    4345    6180
Encroach Node=29340
       1    4345    6180
Encroach Node=29193
       1    5850    7530
Encroach Node=28793
       1    5460    7152
Encroach Node=28133
       1    4878    6832
Encroach Node=27273
       1    4266    6534
Encroach Node=26366
       1    3247    5633
Encroach Node=25273
       1    2827    5465
Encroach Node=24894
       1    2831    5347
Encroach Node=24559
       1    2689    5291
Encroach Node=23599
       1    2000    5027
Encroach Node=22674
       1    1000    4745
Encroach Node=22635
       1    1000    4755
Encroach Node=22564
       1    1100    4779
Encroach Node=22475
       1    1100    4753
Encroach Node=22474
       1    1200    4753
Encroach Node=22381
       1    1500    4681
Encroach Node=21359
       1    1900    4884
Encroach Node=20505
       1    1900    5020
Encroach Node=19503
       1    3000    5139
Encroach Node=18646
       1    3556    5500
Encroach Node=18588
       1    3580    5485
Encroach Node=18587
       1    3596    5498
Encroach Node=18582
       1    3600    5488
Encroach Node=18581
       1    3618    5500
Encroach Node=18546
       1    3700    5500
Encroach Node=17640
       1    1870    3550
Encroach Node=16674
       1    1100    2600
Encroach Node=15704
       1    1096    2493
Encroach Node=14673
       1    1098    2464
Encroach Node=14572
       1    1070    2500
Encroach Node=14570
       1    1047    2479
Encroach Node=14435
       1    1047    2515
Encroach Node=14343
       1    1105    2462
Encroach Node=14088
       1    1105    2460
Encroach Node=13974
       1    1094    2442
Encroach Node=13972
       1    1113    2463
Encroach Node=13953
       1    1114    2476
Encroach Node=13952
       1    1103    2465
Encroach Node=13868
       1    1105    2464
Encroach Node=13319
       1    1083    2471
Encroach Node=12684
       1    1100    2550
Encroach Node=11602
       1    1106    2532
Encroach Node=10558
       1    1111    2492
Encroach Node=9620
       1    1107    2553
Encroach Node=8625
       1    1101    2550
Encroach Node=7854
       1    1105    2464
Encroach Node=7380
       1    1186    2500
Encroach Node=6809
       1    1110    2484
Encroach Node=6715
       1    1050    2500
Encroach Node=6694
       1    1050    2500
Encroach Node=6693
       1    1050    2500
Encroach Node=6689
       1    1050    2500
Encroach Node=6669
       1    1060    2500
Encroach Node=6589
       1    1116    2481
Encroach Node=5991
       1    1125    2461
Encroach Node=5464
       1    1140    2405
Encroach Node=4951
       1    1131    2418
Encroach Node=4851
       1    1033    2500
Encroach Node=4789
       1    1033    2500
Encroach Node=4788
       1    1086    2550
Encroach Node=4679
       1    1159    2498
Encroach Node=4102
       1    1100    2700
Encroach Node=3322
       1    1100    2654
Encroach Node=3211
       1 1029.11  2749.8
Encroach Node=3140
       1 1029.13 2749.78
Encroach Node=3139
       1    1030    2749
Encroach Node=3040
       1    1048    2709
Encroach River=Elm Fork Split1
Encroach Reach=efs1
Encroach Node=9111
       1    1410    3000
Encroach Node=9090
       1    1400    2995
Encroach Node=8953
       1    1150    2840
Encroach Node=8594
       1    1050    2620
Encroach Node=8418
       1    1050    2640
Encroach Node=8287
       1    1050    2800
Encroach Node=8217
       1    1050    2800
Encroach Node=8084
       1    1050    2800
Encroach Node=7856
       1    1050    2970
Encroach Node=7640
       1    1050    3030
Encroach Node=7363
       1    1050    3100
Encroach Node=6926
       1    1050    3055
Encroach Node=6448
       1    1150    3100
Encroach Node=6108
       1    1350    3240
Encroach Node=5842
       1    1341    3250
Encroach Node=5127
       1    1365    3301
Encroach Node=4677
       1    1693    3754
Encroach Node=4346
       1    1611    3463
Encroach Node=4072
       1    1750    3114
Encroach Node=3808
       1    1798    2900
Encroach Node=3526
       1    1720    2800
Encroach Node=3190
       1    1750    2700
Encroach Node=2907
       1    1500    2750
Encroach Node=2515
       1    1444    2531
Encroach Node=2444
       1    1480    2531
Encroach Node=2242
       1    1628    2330
Encroach Node=2036
       1    1600    2330
Encroach Node=1936
       1    1600    2368
Encroach Node=1860
       1    1300    2041
Encroach Node=1527
       1    1370    2111
Encroach Node=1069
       1    1558    2231
Encroach Node=889
       1    1419    2120
Encroach Node=712
       1    1390    1997
Encroach Node=408
       1    1249    1739
Encroach Node=81
       1    1040    1550
Encroach River=Elm Fork L-Spill
Encroach Reach=efl
Encroach Node=15577
       1    1100    1650
Encroach Node=14999
       1    1300    1520
Encroach Node=13559
       1    1330    1512
Encroach Node=12699
       1    1463    1648
Encroach Node=11887
       1    1703    2248
Encroach Node=11867
       1    1703    2248
Encroach Node=11765
       1    1703    2248
Encroach Node=10503
       1    2195    2496
Encroach Node=9797
       1    2105    2400
Encroach Node=9029
       1    1492    1690
Encroach Node=8297
       1    1414    1685
Encroach Node=7346
       1    1482    1828
Encroach Node=7275
       1    1587    1800
Encroach Node=6696
       1    1450    1600
Encroach Node=5924
       1    1753    1970
Encroach Node=5486
       1    1720    1930
Encroach Node=5073
       1    1900    2414
Encroach Node=4421
       1    2220    4200
Encroach Node=3500
       1    1909    3793
Encroach River=Elm Fork Split2
Encroach Reach=efs2
Encroach Node=133117
       1    8920    9472
Encroach Node=132963
       1    8790    9101
Encroach Node=132716
       1    8928    9400
Encroach Node=132009
       1    8896    9850
Encroach Node=131340
       1    9078   10239
Encroach Node=130588
       1    9128   10139
Encroach Node=130020
       1    9051    9771
Encroach Node=129432
       1    9365    9792
Encroach Node=128911
       1    9653   10010
Encroach Node=128358
       1    6057    6552
Encroach Node=127822
       1    4150    4690
Encroach Node=127374
       1    3035    3539
Encroach Node=126920
       1    2419    2825
Encroach Node=126305
       1    1984    2319
Encroach Node=126304
       1    1984    2319
Encroach Node=126185
       1    1867    2223
Encroach Node=126184
       1    1867    2223
Encroach River=Main Stem
Encroach Reach=ms
Encroach Node=148139
       1       0    3146
Encroach Node=147967
       1       0    3067
Encroach Node=147799
       1       0    3006
Encroach Node=147633
       1       0    3003
Encroach Node=147473
       1       0    3019
Encroach Node=147285
       1       0    3004
Encroach Node=147100
       1       0    2997
Encroach Node=146913
       1       0    2996
Encroach Node=146727
       1       0    3002
Encroach Node=146534
       1       0    3008
Encroach Node=146346
       1       0    3021
Encroach Node=146157
       1       0    3041
Encroach Node=145971
       1      29    3119
Encroach Node=145772
       1      29    3119
Encroach Node=145578
       1       0    3062
Encroach Node=145385
       1       0    3020
Encroach Node=145198
       1       0    2988
Encroach Node=145017
       1       0    2954
Encroach Node=144841
       1       0    2937
Encroach Node=144664
       1       0    2933
Encroach Node=144488
       1       0    2925
Encroach Node=144317
       1       0    2921
Encroach Node=144130
       1       0    2932
Encroach Node=143948
       1       0    2932
Encroach Node=143766
       1       0    2930
Encroach Node=143584
       1       0    2934
Encroach Node=143406
       1       0    2929
Encroach Node=143213
       1       0    2925
Encroach Node=143026
       1       0    2925
Encroach Node=142839
       1       0    2925
Encroach Node=142657
       1       0    2921
Encroach Node=142436
       1       0    2930
Encroach Node=142221
       1       0    2923
Encroach Node=142005
       1       0    2917
Encroach Node=141794
       1       0    2915
Encroach Node=141578
       1       0    2910
Encroach Node=141367
       1       0    2908
Encroach Node=141156
       1       0    2902
Encroach Node=140944
       1       0    2896
Encroach Node=140844
       1       0    2888
Encroach Node=140738
       1    1000    3902
Encroach Node=140650
       1    1000    3935
Encroach Node=140553
       1    1000    3908
Encroach Node=140453
       1       0    2897
Encroach Node=140272
       1       0    2892
Encroach Node=140096
       1       0    2890
Encroach Node=139921
       1       0    2903
Encroach Node=139745
       1       0    2898
Encroach Node=139574
       1       0    2895
Encroach Node=139379
       1       0    2906
Encroach Node=139189
       1       0    2893
Encroach Node=138999
       1       0    2864
Encroach Node=138814
       1       0    2812
Encroach Node=138618
       1       0    2748
Encroach Node=138427
       1       0    2710
Encroach Node=138236
       1       0    2690
Encroach Node=138050
       1       0    2681
Encroach Node=137821
       1       0    2707
Encroach Node=137598
       1       0    2769
Encroach Node=137374
       1       0    2840
Encroach Node=137150
       1       0    2898
Encroach Node=136930
       1       0    2937
Encroach Node=136719
       1       0    2958
Encroach Node=136513
       1       0    2963
Encroach Node=136308
       1       0    2967
Encroach Node=136103
       1       0    2975
Encroach Node=135903
       1       0    2981
Encroach Node=135709
       1       0    2978
Encroach Node=135519
       1       0    2984
Encroach Node=135329
       1       0    2991
Encroach Node=135139
       1       0    3002
Encroach Node=134953
       1       0    3012
Encroach Node=134884*
       1       7    3020
Encroach Node=134770*
       1       7    3017
Encroach Node=134698
       1       0    3010
Encroach Node=134503
       1       0    2999
Encroach Node=134309
       1       0    2975
Encroach Node=134115
       1       0    2933
Encroach Node=133926
       1       0    2891
Encroach Node=133738
       1       0    2858
Encroach Node=133515
       1       0    2808
Encroach Node=133295
       1       0    2754
Encroach Node=133073
       1       0    2710
Encroach Node=132850
       1       0    2667
Encroach Node=132625
       1       0    2652
Encroach Node=132416
       1       0    2634
Encroach Node=132205
       1       0    2624
Encroach Node=131995
       1       0    2618
Encroach Node=131785
       1       0    2608
Encroach Node=131575
       1       0    2604
Encroach Node=131360
       1       0    2589
Encroach Node=131143
       1       0    2579
Encroach Node=130926
       1       0    2575
Encroach Node=130706
       1       0    2555
Encroach Node=130531
       1       0    2554
Encroach Node=130353
       1       0    2551
Encroach Node=130175
       1       0    2541
Encroach Node=129997
       1       0    2542
Encroach Node=129817
       1       0    2537
Encroach Node=129640
       1       0    2520
Encroach Node=129459
       1       0    2513
Encroach Node=129281
       1       0    2515
Encroach Node=129100
       1       0    2506
Encroach Node=128914
       1       0    2489
Encroach Node=128725
       1       0    2490
Encroach Node=128533
       1       0    2484
Encroach Node=128318
       1     992    3465
Encroach Node=128286
       1     992    3465
Encroach Node=128067
       1       0    2483
Encroach Node=127936
       1   972.5    3444
Encroach Node=127903
       1   972.5    3436
Encroach Node=127722
       1     980    3436
Encroach Node=127692
       1     980    3435
Encroach Node=127495
       1       0    2444
Encroach Node=127288
       1       0    2439
Encroach Node=127100
       1       0    2441
Encroach Node=126920
       1       0    2424
Encroach Node=126738
       1       0    2414
Encroach Node=126556
       1       0    2410
Encroach Node=126371
       1       0    2398
Encroach Node=126243
       1       0    2394
Encroach Node=126062
       1       0    2385
Encroach Node=125881
       1       0    2373
Encroach Node=125696
       1       0    2354
Encroach Node=125485
       1       0    2314
Encroach Node=125270
       1       0    2271
Encroach Node=125053
       1       0    2219
Encroach Node=124837
       1       0    2173
Encroach Node=124615
       1       0    2127
Encroach Node=124432
       1       0    2078
Encroach Node=124240
       1       0    2013
Encroach Node=124048
       1       0    1975
Encroach Node=123848
       1       0    1952
Encroach Node=123657
       1       0    1940
Encroach Node=123499
       1       0    1932
Encroach Node=123430
       1       0    1933
Encroach Node=123337
       1       0    1933
Encroach Node=123157
       1       0    1922
Encroach Node=122948
       1       0    1940
Encroach Node=122886
       1    1000    2972
Encroach Node=122833
       1    1000    2970
Encroach Node=122747
       1       0    1920
Encroach Node=122553
       1    1009    2920
Encroach Node=122429
       1    1009    2920
Encroach Node=122374
       1       0    1913
Encroach Node=122192
       1       0    1949
Encroach Node=122038
       1       0    1977
Encroach Node=121877
       1       0    2001
Encroach Node=121707
       1       0    2054
Encroach Node=121623
       1    1000    3082
Encroach Node=121591
       1    1000    3081
Encroach Node=121501
       1       0    2019
Encroach Node=121344
       1       0    1934
Encroach Node=121174
       1       0    1859
Encroach Node=121002
       1       0    1850
Encroach Node=120814
       1       0    1868
Encroach Node=120764
       1    1021    2918
Encroach Node=120688
       1    1000    2905
Encroach Node=120613
       1       0    1915
Encroach Node=120481
       1       0    1883
Encroach Node=120335
       1       0    1915
Encroach Node=120175
       1       0    1927
Encroach Node=120017
       1       0    1931
Encroach Node=119848
       1       0    1928
Encroach Node=119681
       1       0    1925
Encroach Node=119501
       1       0    1919
Encroach Node=119331
       1       0    1916
Encroach Node=119146
       1       0    1929
Encroach Node=118962
       1       0    1931
Encroach Node=118766
       1       0    1937
Encroach Node=118699
       1    1037    2979
Encroach Node=118603
       1    1000    2942
Encroach Node=118516
       1       0    1940
Encroach Node=118366
       1       0    1948
Encroach Node=118280
       1       0    1953
Encroach Node=118063
       1       0    1957
Encroach Node=117983
       1       0    1949
Encroach Node=117909
       1       0    1944
Encroach Node=117797
       1       0    1933
Encroach Node=117660
       1       0    1923
Encroach Node=117560
       1       0    1914
Encroach Node=117392
       1       0    1907
Encroach Node=117282
       1       0    1911
Encroach Node=117114
       1       0    1918
Encroach Node=116938
       1       0    1921
Encroach Node=116758
       1       0    1927
Encroach Node=116611
       1       0    1925
Encroach Node=116461
       1       0    1923
Encroach Node=116305
       1       0    1930
Encroach Node=116233
       1    1006    2961
Encroach Node=116174
       1     997    2988
Encroach Node=116101
       1       0    1954
Encroach Node=115932
       1       0    1907
Encroach Node=115756
       1     -56    1845
Encroach Node=115697
       1     -63    1831
Encroach Node=115625
       1       0    1884
Encroach Node=115432
       1       0    1865
Encroach Node=115234
       1       0    1863
Encroach Node=115029
       1       0    1867
Encroach Node=114895
       1       0    1874
Encroach Node=114762
       1       0    1900
Encroach Node=114634
       1       0    1962
Encroach Node=114564
       1      52    2027
Encroach Node=114502
       1      32    2018
Encroach Node=114449
       1       0    1984
Encroach Node=114232
       1       0    1924
Encroach Node=114186
       1      14    1900
Encroach Node=114110
       1       0    1915
Encroach Node=114044
       1       0    1910
Encroach Node=113886
       1       0    1917
Encroach Node=113722
       1       0    1933
Encroach Node=113551
       1       0    1942
Encroach Node=113398
       1       0    1969
Encroach Node=113240
       1       0    1998
Encroach Node=113083
       1       0    2025
Encroach Node=112922
       1       0    2065
Encroach Node=112872
       1       0    2053
Encroach Node=112772
       1       0    2077
Encroach Node=112627
       1       0    2093
Encroach Node=112467
       1       0    2097
Encroach Node=112302
       1       0    2090
Encroach Node=112124
       1       0    2066
Encroach Node=111937
       1       0    1991
Encroach Node=111742
       1       0    1919
Encroach Node=111569
       1       0    1876
Encroach Node=111392
       1       0    1884
Encroach Node=111212
       1       0    1904
Encroach Node=111064
       1       0    1918
Encroach Node=110918
       1       0    1945
Encroach Node=110773
       1       0    1977
Encroach Node=110615
       1       0    2022
Encroach Node=110460
       1       0    2081
Encroach Node=110332
       1       0    2123
Encroach Node=110205
       1       0    2172
Encroach Node=110079
       1       0    2239
Encroach Node=110001
       1    1002    3275
Encroach Node=109948
       1    1002    3299
Encroach Node=109873
       1       0    2333
Encroach Node=109660
       1       0    2420
Encroach Node=109447
       1       0    2575
Encroach Node=109234
       1       0    2753
Encroach Node=109023
       1       0    2920
Encroach Node=108856
       1       0    2895
Encroach Node=108851
       1       0    2890
Encroach Node=108679
       1       0    2845
Encroach Node=108675
       1       0    2835
Encroach Node=108543*
       1     890    3710
Encroach Node=108521
       1    1024    3840
Encroach Node=108504
       1    1009    3826
Encroach Node=108446*
       1     956    3788
Encroach Node=108361
       1     890    3810
Encroach Node=108328
       1     890    3840
Encroach Node=108289
       1     940    3950
Encroach Node=108267
       1     940    3950
Encroach Node=108261
       1     940    3950
Encroach Node=108242*
       1    1095    4120
Encroach Node=108231
       1    1182    4195
Encroach Node=108150*
       1    1807    4911
Encroach Node=108120
       1    2040    5000
Encroach Node=108107
       1    2072    5000
Encroach Node=108091*
       1    2116    5034
Encroach Node=107955
       1    2480    5350
Encroach Node=107769
       1    1980    4800
Encroach Node=107764
       1    1980    4800
Encroach Node=107547
       1    3165    6000
Encroach Node=107542
       1    3165    6000
Encroach Node=107123
       1    1000    3775
Encroach Node=106645
       1    1000    3600
Encroach Node=106109
       1    1000    3600
Encroach Node=105392
       1    1000    3630
Encroach Node=105323
       1    1000    3610
Encroach Node=104947
       1     800    3523
Encroach Node=104451
       1     700    3528
Encroach Node=103950
       1     600    3610
Encroach Node=103525
       1     100    3550
Encroach Node=103445
       1     150    3550
Encroach Node=102784
       1     750    3950
Encroach Node=101784
       1     800    3920
Encroach Node=101135
       1    1000    3637
Encroach Node=100444
       1    1010    3560
Encroach Node=99788
       1    1010    3500
Encroach Node=99143
       1    1000    3562
Encroach Node=98639
       1    1010    3618
Encroach Node=98178
       1    1010    3585
Encroach Node=97719
       1    1010    3560
Encroach Node=97266
       1    1010    3520
Encroach Node=97059
       1    1010 3541.06
Encroach Node=96783
       1    1040    3560
Encroach Node=96632
       1    1011    3580
Encroach Node=96582
       1    1041    3608
Encroach Node=96331
       1    1061    3559
Encroach Node=96276
       1    1010    3520
Encroach Node=95753
       1    1010    3287
Encroach Node=95392
       1    1010    3160
Encroach Node=94721
       1    1010    3260
Encroach Node=91399
       1    1010    3811
Encroach Node=90942
       1    1010    3890
Encroach Node=90547
       1    1010    3819
Encroach Node=90463
       1    1104    3771
Encroach Node=90224
       1    1036    3955
Encroach Node=90006
       1    1010    4080
Encroach Node=89746
       1    1010    4150
Encroach Node=89539
       1    1010    4103
Encroach Node=89510
       1    1010    4103
Encroach Node=89093
       1    1010    4580
Encroach Node=88616
       1    4854    9656
Encroach Node=87328
       1   14520   19800
Encroach Node=85914
       1   13608   21769
Encroach Node=84656
       1   10200   20384
Encroach Node=83381
       1   10182   18710
Encroach Node=82348
       1    1644    7526
Encroach Node=81776
       1    2478    7775
Encroach Node=81193
       1    3185    8371
Encroach Node=80625
       1    3517    8910
Encroach Node=80021
       1    3850    8700
Encroach Node=79333
       1    3600    8590
Encroach Node=78595
       1    3500    8358
Encroach Node=77823
       1    3500    8252
Encroach Node=76808
       1    3500    7822
Encroach Node=75959
       1    3775    7820
Encroach Node=75877
       1    3775    7820
Encroach Node=75846
       1    3775    7820
Encroach Node=75811
       1    3775    7820
Encroach Node=75196
       1    2800    8330
Encroach Node=74132
       1    2000    8000
Encroach Node=73001
       1    2000    8875
Encroach Node=71491
       1    1923    9039
Encroach Node=69919
       1    2400    9380
Encroach Node=69766
       1    2450    9321
Encroach Node=69176
       1    1600    8158
Encroach Node=68160
       1    2000    8126
Encroach Node=68010
       1    2000    8082
Encroach Node=66412
       1    1118    6249
Encroach Node=63968
       1    1018    6180
Encroach Node=62084
       1     914    5941
Encroach Node=60946
       1    1221    6195
Encroach Node=59442
       1    1072    6228
Encroach Node=58569
       1    1038    6446
Encroach Node=56725
       1    1150    6066
Encroach Node=55873
       1     240    5796
Encroach Node=54986
       1    1277    7204
Encroach Node=53997
       1    1527    8281
Encroach Node=53576
       1     165    6592
Encroach Node=53441
       1     330    6588
Encroach Node=53017
       1    1150    7500
Encroach Node=51999
       1    1156    6882
Encroach Node=51043
       1    1144    6887
Encroach Node=50076
       1    3081    5468
Encroach Node=49896
       1    3080    5455
Encroach Node=48781
       1    1102    6500
Encroach Node=44208
       1    1158    6500
Encroach Node=42574
       1     974    6780
Encroach Node=40237
       1    1058    6780
Encroach Node=37746
       1    1204    7311
Encroach Node=36505
       1    1109    7361
Encroach Node=35176
       1    1060    7427
Encroach Node=32858
       1   10341   16480
Encroach Node=32798
       1   10755   16957
Encroach Node=32751
       1   10755   16957
Encroach Node=32649
       1   10755   16950
Encroach Node=30150
       1   11325   16297
Encroach Node=28996
       1   12258   17152
Encroach Node=27414
       1   11911   16937
Encroach Node=25457
       1    1122    5898
Encroach River=West Fork
Encroach Reach=wf3
Encroach Node=206158
       1    1710 4914.25
Encroach Node=205180
       1    3803    6035
Encroach Node=204260
       1    1230 2962.25
Encroach Node=202984
       1    1085    3005
Encroach Node=200958
       1     956    2850
Encroach Node=199766
       1    1400    3260
Encroach Node=198506
       1    1520    3450
Encroach Node=198115
       1    2396    4140
Encroach Node=197858*
       1    2546    4330
Encroach Node=197618*
       1    2698    4450
Encroach Node=197400*
       1    2849    4560
Encroach Node=197202
       1    3000    4740
Encroach Node=196621
       1    3720    5360
Encroach Node=196275*
       1    4070    5710
Encroach Node=195795*
       1    4110    5800
Encroach Node=195470
       1    4410    6100
Encroach Node=195036
       1    4738    6785
Encroach Node=193898
       1    4280    7284
Encroach Node=193493
       1    3330    6162
Encroach Node=193389
       1    3485    6380
Encroach Node=193310
       1    3446    6409
Encroach Node=193137
       1    3357    6432
Encroach Node=193094
       1    3340    6509
Encroach Node=193034
       1    3410    6623
Encroach Node=192957
       1    3310    6638
Encroach Node=192700
       1    3135    6564
Encroach Node=191569
       1    3292    6794
Encroach Node=191228
       1    3345    6930
Encroach Node=190795
       1    3389    7225
Encroach Node=190401
       1    3390    6910
Encroach Node=190220
       1    3390    6860
Encroach Node=190059
       1    3389    6810
Encroach Node=189845
       1    3392    6825
Encroach Node=189043
       1    3396    6475
Encroach Node=188186
       1    3438    6094
Encroach Node=187587
       1    3652    5630
Encroach Node=187069
       1    4161    5595
Encroach Node=187026
       1    4167    5572
Encroach Node=187022
       1    4167    5572
Encroach Node=187021
       1    3079    4477
Encroach Node=186977
       1    5135    6505
Encroach Node=186799
       1    3120    4352
Encroach Node=186596
       1    2780    4214
Encroach Node=185854
       1    3750    5727
Encroach Node=185333
       1    5420    7046
Encroach Node=184797
       1    6010    7010
Encroach Node=184441
       1 6320.88    6990
Encroach Node=183656
       1    6848    7241
Encroach Node=183043
       1    6925    7307
Encroach Node=182093
       1    6870    7317
Encroach Node=181468
       1    7356    7761
Encroach Node=181426
       1    7424    7814
Encroach Node=181422
       1    7424    7814
Encroach Node=181418
       1    7424    7814
Encroach Node=181314
       1 7481.43 7863.43
Encroach Node=181232
       1 7481.43 7863.43
Encroach Node=181212
       1 7477.91    8030
Encroach Node=180404
       1    7577    8904
Encroach Node=179021
       1    7760    9380
Encroach Node=178611
       1    7820    9600
Encroach Node=178426
       1    1008    2844
Encroach Node=178323
       1    1008    2844
Encroach Node=178206
       1    7650    9580
Encroach Node=177430
       1    7560    9350
Encroach Node=176262
       1    7540    9270
Encroach Node=171852
       1    5410    8520
Encroach Node=165197
       1    5000    8260
Encroach Node=162387
       1    6150    8350
Encroach Node=161687
       1    6360    8525
Encroach Node=161585
       1    6387    8550
Encroach Node=161274
       1  5336.5    7660
Encroach Node=161012
       1    5320    7740
Encroach Node=160831
       1    6330    8670
Encroach Node=160768
       1    6300    8703
Encroach Node=158611
       1    5540    8570
Encroach Node=158504
       1    5720    8800
Encroach Node=158015
       1    6350    9740
Encroach Node=155669
       1    6401    9545
Encroach Node=154482
       1    6480    9650
Encroach Node=154399
       1    6460    9720
Encroach Node=154398
       1    6460    9720
Encroach Node=154357
       1    6460    9720
Encroach Node=154356
       1    6440    9720
Encroach Node=154255
       1    6325    9720
Encroach Node=153249
       1    5850    9720
Encroach Node=151887
       1    6455   11660
Encroach Node=151089
       1    5880   12150
Encroach Node=150329
       1    5350   12280
Encroach Node=149159
       1    4575   12370
Encroach Node=148620
       1 3478.82   12167
Encroach Node=148063
       1    2725 12009.8
Encroach Node=147468
       1    1650 12297.9
Encroach Node=147459
       1    1650 12297.9
Encroach Node=147417
       1    1650 12297.9
Encroach Node=147372
       1    1650 12297.9
Encroach Node=147366
       1    1650 12297.9
Encroach Node=147309
       1    1650 12297.9
Encroach Node=147299
       1    1650 12297.9
Encroach Node=144438
       1  1024.7   13630
Encroach Node=142627
       1  1026.2   12950
Encroach Node=140843
       1  3650.4   13715
Encroach Node=138168
       1    3352   12295
Encroach Node=136890
       1    3463   12370
Encroach Node=133675
       1    2335   10980
Encroach Node=133662
       1    2335   10978
Encroach Node=133505
       1 2146.73   10817
Encroach Node=133461
       1    3088   11788
Encroach Node=133374
       1    3088   11788
Encroach Node=133373
       1    3039 11733.2
Encroach Node=133330
       1    3229 11913.2
Encroach Node=133329
       1    3101 11780.6
Encroach Node=133251
       1    3001 11687.6
Encroach Node=131430
       1    2892   11000
Encroach Node=130880
       1    2892   10290
Encroach Node=130370
       1    2892   10200
Encroach Node=127957
       1  2808.2   10006
Encroach Node=127946
       1  2828.2   10070
Encroach Node=127859
       1  2860.2   10084
Encroach Node=127847
       1  2808.2   10028
Encroach Node=127834
       1  2808.2   10048
Encroach Node=127826
       1  2808.2   10048
Encroach Node=127767
       1  2808.2   10048
Encroach Node=126554
       1    1300    6839
Encroach Node=126526
       1    1300    6839
Encroach Node=126359
       1    1460    6765
Encroach Node=126177
       1    1610  6649.4
Encroach Node=125975
       1    1750  6568.1
Encroach Node=125699
       1    1850  6374.2
Encroach Node=125659
       1     940  5356.3
Encroach Node=125524
       1  1827.7  6287.7
Encroach Node=125234
       1  1916.6    6098
Encroach Node=124978
       1    1994    5909
Encroach Node=124562
       1 2222.82    5788
Encroach Node=124060
       1    2509  5593.5
Encroach Node=123707
       1    2493  5548.5
Encroach Node=123399
       1    2518  5623.2
Encroach Node=123104
       1    2544    5666
Encroach Node=122822
       1    2640  5731.1
Encroach Node=122537
       1  2758.5  5824.1
Encroach Node=122267
       1  2913.2  5923.7
Encroach Node=121845
       1  3107.9  6128.5
Encroach Node=121365
       1    3370  6351.5
Encroach Node=120895
       1 3615.12  6369.8
Encroach Node=120394
       1  4099.8  6658.4
Encroach Node=119702
       1 4118.51    6220
Encroach Node=118850
       1 4349.93    6444
Encroach Node=118334
       1 4564.62    6490
Encroach Node=118069
       1  4662.9    6531
Encroach Node=116629
       1    4550    7020
Encroach Node=116017
       1    4950    8200
Encroach Node=112524
       1    5250    8320
Encroach Reach=wf3f
Encroach Node=112687
       1    5605    7155
Encroach Node=112151
       1    5460    6732
Encroach Node=112054
       1    5760    6760
Encroach Node=111837
       1    5793    6700
Encroach Node=111563
       1    5871    6723
Encroach Node=111531
       1 5906.06 6663.92
Encroach Node=111402
       1 5906.06 6663.92
Encroach Node=111382
       1    5884    6664
Encroach Node=111268
       1    3057    3883
Encroach Node=111043
       1    2836    3764
Encroach Node=110718
       1    2759    3758
Encroach Node=110419
       1    2836    3938
Encroach Node=110041
       1    3018    4211
Encroach Node=109064
       1    3208    4544
Encroach Reach=wf3e
Encroach Node=111697
       1    7155    8550
Encroach Node=111315
       1    8300    9240
Encroach Node=111310
       1    8300    9240
Encroach Node=111296
       1    8300    9240
Encroach Node=111285
       1    8300    9240
Encroach Node=110511
       1    8280    9164
Encroach Node=110200
       1    8800    9430
Encroach Node=109675
       1    9340    9670
Encroach Node=109561
       1    9285    9620
Encroach Node=109482
       1    9379    9624
Encroach Node=109377
       1    9379    9624
Encroach Node=109354
       1    9379    9624
Encroach Node=109186
       1    6470    6719
Encroach Node=108974
       1    6370    6710
Encroach Node=108657
       1    5990    6542
Encroach Node=108546
       1    5634    6390
Encroach Node=108432
       1    5541    6390
Encroach Node=108310
       1    5497    6470
Encroach Node=108049
       1    5384    6480
Encroach Reach=wf3d
Encroach Node=107732
       1    3580    6805
Encroach Node=107216
       1    4077    6848
Encroach Node=106864
       1    4250    7290
Encroach Node=104794
       1    4178    8380
Encroach Node=103963
       1    4530    8820
Encroach Node=102846
       1    4970    9299
Encroach Node=101470
       1    5660    9580
Encroach Node=99962
       1    5485    9345
Encroach Node=99952
       1    5485    9345
Encroach Node=99892
       1    5485    9345
Encroach Node=99886
       1    5485    9345
Encroach Node=97849
       1    5550    8707
Encroach Node=96881
       1    5545 7960.82
Encroach Node=96518
       1    5560    8265
Encroach Node=96217
       1    5400    8200
Encroach Node=96041
       1    5400    8300
Encroach Node=95724
       1    5335    8488
Encroach Node=94344
       1    3744    7450
Encroach Node=92613
       1    3950    7770
Encroach Node=91597
       1    3500    7420
Encroach Node=89818
       1    3232    7347
Encroach Node=88588
       1    3350    7196
Encroach Node=88020
       1    2693    6215
Encroach Node=87403
       1    2249    5730
Encroach Node=86258
       1    2210    5605
Encroach Node=85778
       1    2470    6215
Encroach Reach=wf3b
Encroach Node=84526
       1    1540    4227
Encroach Node=83812
       1    1620    4384
Encroach Node=81994
       1    1780    3184
Encroach Node=81108
       1    2219 2895.44
Encroach Node=80982
       1    2500    2908
Encroach Node=80981
       1    2500    2908
Encroach Node=80891
       1    2500    2908
Encroach Node=80890
       1    2500    2908
Encroach Node=80794
       1    2470    3000
Encroach Node=78277
       1    1929    3421
Encroach Node=78173
       1    2246    3590
Encroach Node=78172
       1    2234    3590
Encroach Node=78162
       1    2240    3590
Encroach Node=78161
       1    2246    3590
Encroach Node=78060
       1    1915    3302
Encroach Reach=wf3c
Encroach Node=80116
       1    4500    5681
Encroach Node=79747
       1    5365    6348
Encroach Node=79496
       1    5163    5985
Encroach Node=79116
       1    5600    6100
Encroach Node=79022
       1    5760    6146
Encroach Node=79008
       1  5756.5  6149.5
Encroach Node=78897
       1    5760    6153
Encroach Node=78886
       1    5760    6153
Encroach Node=78766
       1    5755    6237
Encroach Node=78525
       1    5200    5786
Encroach Node=78408
       1    5300    5705
Encroach Node=78407
       1    5300    5705
Encroach Node=78396
       1    5300    5705
Encroach Node=78394
       1    5300    5705
Encroach Node=78309
       1    4930    5398
Encroach Reach=wf3a
Encroach Node=74827
       1    1270    3642
Encroach Node=73613
       1    1609    3226
Encroach Node=73281
       1    1689    3300
Encroach Node=72546
       1    1867    3605
Encroach Node=72425
       1    1867    3605
Encroach Node=71998*
       1    1580    3285
Encroach Node=71628
       1    1245    3105
Encroach Node=71225
       1    1147    3186
Encroach Node=70832
       1    1365    3425
Encroach Node=69985
       1    1397    3417
Encroach Node=69757
       1    1356    3431
Encroach Node=69168
       1    2760    4587
Encroach Node=68310
       1  2940.8    4490
Encroach Node=67946
       1    2850    4337
Encroach Node=67523
       1    2600  4069.3
Encroach Node=66492
       1    2428    3822
Encroach Node=66018
       1    2453 3733.61
Encroach Node=65487
       1    2453    3589
Encroach Node=63489
       1    2495    3969
Encroach Node=61326
       1    2520    4300
Encroach Node=61222
       1    2570    4300
Encroach Node=61221
       1    2200 3943.47
Encroach Node=61141
       1    2230 3942.66
Encroach Node=61140
       1    2200    3989
Encroach Node=61036
       1    2200    3989
Encroach Node=60462
       1    3250    5173
Encroach Node=59661
       1    3825    5960
Encroach Node=58321
       1    4161    7515
Encroach Node=57570
       1    5910    8890
Encroach Node=57287
       1    5910    8890
Encroach Node=57083
       1    6642    9531
Encroach Node=55744
       1    9441   12251
Encroach Reach=wf2
Encroach Node=53716
       110052.29   12502
Encroach Node=52598
       1   10811 12916.2
Encroach Node=52587
       1   10811 12916.2
Encroach Node=51567
       1   11203   13240
Encroach Node=51466
       1   11203   13240
Encroach Node=50231
       1   11760   13990
Encroach Node=50220
       1   11760   13990
Encroach Node=49464
       1   12774   14700
Encroach Node=48418
       1   13632   15140
Encroach Node=47252
       1   13021   15576
Encroach Node=46316
       1   13058   15515
Encroach Node=45304
       1    7391    9873
Encroach Node=44415
       1   13927   16389
Encroach Node=44332
       1   13040   15423
Encroach Node=44216
       1   13040   15423
Encroach Node=44141
       1   13954   16450
Encroach Node=43868
       1     620    2637
Encroach Node=43719
       1     764    2608
Encroach Node=43418
       1   11847   13630
Encroach Node=42949
       1   11754   13565
Encroach Node=42739
       1   11839   13664
Encroach Node=42318
       1     420    2128
Encroach Node=42238
       1     259    2032
Encroach Node=42111
       1     375    2176
Encroach Node=41686
       1   11825   13787
Encroach Node=40803
       1    3200    5455
Encroach Node=39099
       1    1044    3395
Encroach Node=38863
       1     134    2595
Encroach Node=38799
       1      57    2508
Encroach Node=38599
       1     141    2816
Encroach Node=38434
       1     139    3180
Encroach Node=38198
       1      55    3289
Encroach Node=38103
       1   10052   13361
Encroach Node=38064
       1     120 3557.09
Encroach Node=37855
       1  8293.5   12650
Encroach Node=37004
       1    7861   12296
Encroach Node=35195
       1    7560   11798
Encroach Reach=wf1
Encroach Node=34256
       1    2367    9150
Encroach Node=33352
       1    6770   12430
Encroach Node=33324
       1    2000    7500
Encroach Node=33301
       1    2050    7475
Encroach Node=33288
       1    2100    7450
Encroach Node=33269
       1    2150    7425
Encroach Node=33230
       1    2175    7400
Encroach Node=33191
       1    2210    7375
Encroach Node=33138
       1    2230    7350
Encroach Node=33049
       1    2253    7325
Encroach Node=33000
       1    2253    7300
Encroach Node=32954
       1    7542   12590
Encroach Node=32913
       1    2253    7315
Encroach Node=32766
       1    2300    7270
Encroach Node=32663
       1    2350    7220
Encroach Node=32035
       1    7809   11715
Encroach Node=30626
       1    6600   10327
Encroach Node=29236
       1    6810    9870
Encroach Node=28846
       1    6918    9779
Encroach Node=28726
       1    6918    9778
Encroach Node=28462
       1    6640   10360
Encroach Node=27892
       1    6400   10250
Encroach Node=25427
       1    6250   10040
Encroach Node=24876
       1    4800    8960
Encroach Node=19918
       1    3710    9231
Encroach Node=18819
       1    3860    9597
Encroach Node=18136
       1    2420    8126
Encroach Node=17722
       1    4350    9770
Encroach Node=17512
       1    4300    9650
Encroach Node=16451
       1    3800    8099
Encroach Node=15777
       1    3210    7364
Encroach Node=15050
       1    3335    7314
Encroach Node=14332
       1    2860    6280
Encroach Node=13520
       1    4400    7960
Encroach Node=12809
       1    4205    8040
Encroach Node=11909
       1    3470    7629
Encroach Node=11272
       1    3280    7322
Encroach Node=10678
       1    2725    6964
Encroach Node=10278
       1    4147    8364
Encroach Node=9859
       1    3730    8030
Encroach Node=9764
       1    3850    8000
Encroach Node=9763
       1    2752    6917
Encroach Node=9619
       1    2722    6917
Encroach Node=9618
       1    3810    8000
Encroach Node=9516
       1    3810    8000
Encroach Node=8892
       1    2450    6770
Encroach Node=8489
       1    2465    6737
Encroach Node=8367
       1    2487    6773
Encroach Node=8147
       1    3178    7763
Encroach Node=5786
       1    2885    6345
Encroach Node=4670
       1    3215    6342
Encroach Node=3830
       1    2160    4550
Encroach Node=3323
       1    1890    3760
Encroach Node=2686
       1    1750    3450
Encroach Node=2207
       1    1616    3553
Encroach Node=1494
       1    1435    3747
Encroach River=West Fork Split
Encroach Reach=wfs
Encroach Node=56034
       1      90    1210
Encroach Node=55860
       1  353.25 1138.72
Encroach Node=55343
       1 1738.63 2664.56
Encroach Node=55018
       1 7406.68 8926.64
Encroach Node=54594
       1 5690.93 8015.13
Encroach Node=53266
       1 3980.97 6307.16
Encroach Node=52220
       1 3911.66 5981.64
Encroach Node=51150
       1 2725.88 4547.18
Encroach Node=50291
       1 2594.29 4227.93
Encroach Node=49493
       1    5658    6158
Encroach Node=48553
       1    5757    6007
Encroach Node=48383
       1    5797    5937
Encroach Node=48280
       1    6630    7290
Encroach Node=48075
       1    5600    6410
Encroach Node=47579
       1 4259.81  6059.3
Encroach Node=46993
       1  993.72 3720.52
Encroach Node=46031
       1 1400.84 3732.74
Encroach Node=44904
       1 2306.98 3805.72
Encroach Node=40891
       1 1394.74 2426.75
Encroach Node=40604
       1    1224    2408
Encroach Node=40508*
       1 1337.81 2535.61
Encroach Node=40505
       1  1348.5 2674.86
Encroach Node=40500
       1 1309.86 2782.51
Encroach Node=40485
       1 1220.87 2703.53
Encroach Node=40479
       1 1364.13 2860.24
Encroach Node=40362
       1    1400    3060
Encroach Node=39084
       1     184    2290
Encroach Node=38783
       1    5867    8007
Flow Ratio Tolerance=0.1
Flow Ratio Min Ratio=0.5
Flow Ratio Max Ratio=4
Flow Ratio Max Iterations= 10
BEGIN DESCRIPTION:
Existing Model
This plan is valid downstream of West Fork cross-section 206218 for the West Fork, Elm Fork, and Trinity River Main Stem.  This plan represents the FEMA Floodway using the 1% AEP peak flows and the NFIP 10%, 4%, 2%, 1% geometry.
END DESCRIPTION:
Computation Interval=1HOUR
Output Interval=1HOUR
Instantaneous Interval=1HOUR
Mapping Interval=1HOUR
Computation Time Step Use Courant=        0
Computation Time Step Use Time Series=    0
Computation Time Step Count To Double=0
Computation Time Step Max Doubling=0
Computation Time Step Max Halving=0
Computation Time Step Residence Courant=0
Run HTab= 0
Run UNet= 0
Run Sediment= 0
Run PostProcess= 0
Run WQNet= 0
Run RASMapper= 0
UNET Theta= 1
UNET Theta Warmup= 1
UNET ZTol= 0.02
UNET ZSATol= 0.05
UNET MxIter= 20
UNET Max Iter WO Improvement= 0
UNET MaxInSteps= 0
UNET DtIC= 0
UNET DtMin= 0
UNET MaxCRTS= 20
UNET WFStab= 2
UNET SFStab= 1
UNET WFX= 1
UNET SFX= 1
UNET Gravity=32.17405
UNET 1D Methodology=Finite Difference
UNET DSS MLevel= 4
UNET Pardiso=0
UNET DZMax Abort= 100
UNET Use Existing IB Tables=-1
UNET Froude Reduction=False
UNET Froude Limit= 1
UNET Froude Power= 10
UNET D1 Cores= 0
UNET WindReference=Eulerian
UNET WindDragFormulation=Hsu (1988)
UNET D2 Coriolis=0
UNET D2 Cores= 0
UNET D2 Theta= 1
UNET D2 Theta Warmup= 1
UNET D2 Z Tol= 0.01
UNET D2 Volume Tol= 0.01
UNET D2 Max Iterations= 20
UNET D2 Advanced Convergence=0
UNET D2 WS Max Tol=0.15
UNET D2 WS RMS Tol=0.002
UNET D2 WS Stall Tol=1
UNET D2 Equation= 0
UNET D2 RampUpFraction=0.1
UNET D2 TimeSlices= 1
UNET D2 Turbulence Formulation=Non-Conservative (original)
UNET D2 Eddy Viscosity=0.3
UNET D2 Transverse Eddy Viscosity=0.3
UNET D2 Smagorinsky Mixing=0
UNET D2 BCVolumeCheck=0
UNET D2 Cores=0
UNET D2 SolverType=PARDISO (Direct)
UNET D2 Minimum Iterations= 3
UNET D2 Maximum Iterations= 30
UNET D2 Restart Number= 10
UNET D2 Relaxation Coeff=1.3
UNET D2 SOR Precondition Iterations= 10
UNET D2 ILUT Maximum Fill= 8
UNET D2 ILUT Tolerance=1E-08
UNET D2 Convergence Tolerance=0.00001
PS Theta= 1
PS WS Tol= 0.01
PS Volume Tol= 0.01
PS Max Iterations= 20
PS Equation= 0
PS Advance Time Step=-1
PS Target Courant=0.9
PS Time Slices= 1
PS Iterate With 2D=0
PS Project Initial WSE from DS=-1
PS Ramp Up Initial WSE from US=-1
PS Cores=0
UNET D1D2 MaxIter= 0
UNET D1D2 ZTol=0.01
UNET D1D2 QTol=0.1
UNET D1D2 MinQTol=1
DSS File=dss
Write IC File= 0
Write IC File at Fixed DateTime=0
Write IC File at Sim End=0
Echo Input=False
Echo Parameters=False
Echo Output=False
Write Detailed= 0
HDF Write Warmup=0
HDF Write Time Slices=0
HDF Flush=0
HDF Compression= 1
HDF Chunk Size= 1
HDF Spatial Parts= 1
HDF Use Max Rows=0
HDF Fixed Rows= 1
Calibration Method= 0
Calibration Iterations= 20
Calibration Max Change=0.05
Calibration Tolerance=0.2
Calibration Maximum=1.5
Calibration Minimum=0.5
Calibration Optimization Method= 1
WQ AD Non Conservative
WQ ULTIMATE=-1
WQ Max Comp Step=1HOUR
WQ Output Interval=15MIN
WQ Output Selected Increments= 0
WQ Create Restart=0
WQ Fixed Restart=0
WQ System Summary=0
WQ Write To DSS=0
Sorting and Armoring Iterations= 10
XS Update Threshold= 0.02
Bed Roughness Predictor= 0
Processes Affected by Predictor=Sediment Only
Hydraulics Update Threshold= 0.02
Energy Slope Method= 2
Volume Change Method= 0
Sediment Retention Method= 0
Sediment TS Multiplier= 1
Warm Up Method= 0
XS Weighting Method= 0
Number of US Weighted Cross Sections= 1
Number of DS Weighted Cross Sections= 1
Upstream XS Weight=0.25
Main XS Weight=0.5
Downstream XS Weight=0.25
Number of DS XS's Weighted with US Boundary= 1
Upstream Boundary Weight= 1
Weight of XSs Associated with US Boundary= 0
Number of US XS's Weighted with DS Boundary= 1
Downstream Boundary Weight= 0.5
Weight of XSs Associated with DS Boundary= 0.5
Percentile Method= 0
Sediment Output Level= 4
Mass or Volume Output= 0
Output Increment Type= 1
Profile and TS Output Increment= 10
Transport Output Increment 1
XS Output Flag= 0
XS Output Increment= 10
Read HDF5 Sediment Hotstart= 0
Sediment Hotstart Type= 0
Write Gradation File= 0
Read Gradation Hotstart= 0
Write HDF5 File= 1
Write Binary Output= 1
Write DSS Sediment File= 0
DSS Sediment Output Type= 1
SV Curve= 0
Specific Gage Flag= 0
Subcell Erosion Methods= 0
Subcell Deposition Methods= 0
Advection Scheme= 1
Matrix Solver= 0
Implicit Weighting Factor= 1
Maximum Outer Loop Convergence Iterations= 5
Convergence Maximum Absolute= 0.001
Convergence RMSE= 0.0001
Grain Fractions Max Abs Error= 0.001
Max Subgrid Regions= 1
Max Subgrid Length Scale= 3.402823E+38
Initial Layer Thickness= 3
Min Layer Thickness= 0.1
Max Layer Thickness= 6
Number of Layers= 5
