HEC-RAS study CDC_Consolidated_Model.prj: Upper Trinity CDC Consolidated Model

--- CDC_Consolidated_Model.p05 (plan) ---

Plan Title=Exist: FEMA Floodway [WF/CF]
Program Version=6.60
Short Identifier=Existing Plan 5
Geom File=g03
Flow File=f05
Subcritical Flow
K Sum by GR= 0
Std Step Tol= 0.01
Critical Tol= 0.01
Num of Std Step Trials= 20
Max Error Tol= 0.3
Flow Tol Ratio= 0.001
Split Flow NTrial= 30
Split Flow Tol= 0.02
Split Flow Ratio= 0.02
Log Output Level= 0
Friction Slope Method= 1
Unsteady Friction Slope Method= 2
Unsteady Bridges Friction Slope Method= 1
Parabolic Critical Depth
Global Vel Dist= 0 , 0 , 0
Global Log Level= 0
CheckData=True
Encroach Param= 0 ,0,0, 2
Encroach River=Clear Fork
Encroach Reach=cf
Encroach Node=64970
       1 4123.93 4317.75
Encroach Node=64699
       1    4090 4302.81
Encroach Node=63740
       1 3330.41    3541
Encroach Node=62334
       1 2184.87 2330.64
Encroach Node=61786
       1 2494.93 2656.54
Encroach Node=60875
       1 2347.36 2531.26
Encroach Node=59870
       1 2497.75 2665.35
Encroach Node=58305
       1 3874.51  4007.2
Encroach Node=56520
       1    3037    3291
Encroach Node=54327
       1    3863    4114
Encroach Node=53445
       1    3261    3503
Encroach Node=52896
       1    3370    3590
Encroach Node=51792
       1    3316    3734
Encroach Node=51743
       1    3319    3740
Encroach Node=51691
       1    3319    3740
Encroach Node=51188
       1    3154    3311
Encroach Node=50198
       1 2566.19  2687.5
Encroach Node=49033
       1    3020  3164.5
Encroach Node=46371
       1    4511    4657
Encroach Node=46285
       1    1347    1485
Encroach Node=46280
       1    1347    1485
Encroach Node=46178
       1    1347    1485
Encroach Node=46177
       1    1347    1485
Encroach Node=45846
       1    4080    4293
Encroach Node=45214
       1  4081.2  4231.5
Encroach Node=44689
       1    4047  4165.9
Encroach Node=44021
       1    3445    3596
Encroach Node=43004
       1  3396.4 4288.16
Encroach Node=40758
       1  1410.7    2434
Encroach Node=39921
       1    2198  2488.8
Encroach Node=39820
       1    1132    1476
Encroach Node=39717
       1    1132    1476
Encroach Node=39619
       1    2209  2632.9
Encroach Node=39124
       1  1781.1  2046.5
Encroach Node=38847
       1    3488  3751.5
Encroach Node=38788
       1  3500.4  3740.4
Encroach Node=38770
       1  3500.4  3740.3
Encroach Node=38484
       1    3610  3842.3
Encroach Node=37851
       1    3664    3937
Encroach Node=37209
       1    3644    3980
Encroach Node=36226
       1  3500.1    3798
Encroach Node=35730
       1    3256  3510.9
Encroach Node=35316
       1    2804    3086
Encroach Node=34851
       1    2783    3092
Encroach Node=34792
       1    2770    3065
Encroach Node=34732
       1    2757    3054
Encroach Node=34705
       1    2692    2935
Encroach Node=34655
       1    2693    2934
Encroach Node=34639
       1    2608    2846
Encroach Node=34592
       1    2608    2843
Encroach Node=34477
       1 2690.72    2967
Encroach Node=33891
       1    2659    2901
Encroach Node=33357
       1    2813    3054
Encroach Node=32715
       1    1971    2213
Encroach Node=32588
       1    1803    2048
Encroach Node=32567
       1    1777    2021
Encroach Node=32374
       1    1778    2019
Encroach Node=32147
       1    1496    1738
Encroach Node=31544
       1    1173    1419
Encroach Node=30698
       1    1070    1310
Encroach Node=29975
       1    4238    4482
Encroach Node=29468
       1    4335    4578
Encroach Node=29447
       1    4335    4578
Encroach Node=29422
       1    4336    4576
Encroach Node=29347
       1    4324    4559
Encroach Node=29295
       1    4324    4559
Encroach Node=29247
       1    4325    4558
Encroach Node=28511
       1    4049    4283
Encroach Node=27187
       1    3629    3870
Encroach Node=26124
       1    2848    3095
Encroach Node=25576
       1    2361    2615
Encroach Node=25574
       1    2361  2614.9
Encroach Node=25532
       1    2302    2558
Encroach Node=25451
       1    2212    2468
Encroach Node=25409
       1  2160.1    2418
Encroach Node=25408
       1  2160.1    2418
Encroach Node=25246
       1    2049    2308
Encroach Node=25146
       1    1988    2239
Encroach Node=24285
       1    1588    1841
Encroach Node=24183
       1    1420    1677
Encroach Node=24119
       1    1592 1848.73
Encroach Node=24025
       1    1611  1860.2
Encroach Node=23921
       1    1621 1875.82
Encroach Node=23362
       1    1552    1796
Encroach Node=22435
       1    1305    1554
Encroach Node=21678
       1    1350    1604
Encroach Node=21161
       1    1382    1642
Encroach Node=21111
       1    1382    1643
Encroach Node=21061
       1    1383    1641
Encroach Node=20182
       1    1466    1737
Encroach Node=19478
       1    1527  1797.9
Encroach Node=18718
       1  1910.4  2168.7
Encroach Node=18134
       1  2322.8  2594.2
Encroach Node=17609
       1  2462.1    2767
Encroach Node=17561*
       1    2480    2781
Encroach Node=17512*
       1  2497.1    2795
Encroach Node=17464*
       1    2515    2814
Encroach Node=17416*
       1    2532  2822.8
Encroach Node=17368*
       1    2550    2836
Encroach Node=17320*
       1    2567    2850
Encroach Node=17271*
       1    2585    2864
Encroach Node=17222*
       1    2595  2877.9
Encroach Node=17173
       1    2618    2891
Encroach Node=17124*
       1    2674    2952
Encroach Node=17075
       1    2729    3012
Encroach Node=17031
       1    2729    3012
Encroach Node=16996.3*
       1    2757    3029
Encroach Node=16961.6*
       1    2784    3045
Encroach Node=16927
       1    2813    3062
Encroach Node=16882.7*
       1    2802    3063
Encroach Node=16838.4*
       1    2792    3064
Encroach Node=16794.1*
       1    2782    3065
Encroach Node=16749.8*
       1    2772    3065
Encroach Node=16705.5*
       1    2763    3066
Encroach Node=16661.2*
       1    2755    3066
Encroach Node=16617
       1  2758.1    3066
Encroach Node=16568*
       1    2830    3140
Encroach Node=16518*
       1    2914  3213.8
Encroach Node=16468*
       1    3000    3286
Encroach Node=16419
       1    3087    3358
Encroach Node=16371*
       1    3054  3338.9
Encroach Node=16324*
       1    3022    3321
Encroach Node=16278*
       1 2990.15  3299.5
Encroach Node=16231*
       1    2959 3277.67
Encroach Node=16185*
       1    2927    3255
Encroach Node=16138
       1    2895    3234
Encroach Node=16103*
       1    2890    3236
Encroach Node=16067*
       1    2908    3238
Encroach Node=16031
       1    2914    3240
Encroach Node=15989
       1    2914    3240
Encroach Node=15970
       1    2902    3266
Encroach Node=15923
       1    2902    3266
Encroach Node=15886.3*
       1    2927    3319
Encroach Node=15849.6*
       1    2961    3373
Encroach Node=15813
       1  2995.2  3422.9
Encroach Node=15479
       1 1024.55    1304
Encroach Node=15323
       1  1026.3    1303
Encroach Node=14832
       1  1026.5    1306
Encroach Node=14181
       1 1022.21    1306
Encroach Node=13358
       1 1201.43 1471.71
Encroach Node=13297
       1 1201.62 1471.55
Encroach Node=13150
       1 1200.68    1470
Encroach Node=12958
       1 1307.42    1510
Encroach Node=12830
       1 1305.16    1558
Encroach Node=12698
       1 1305.16    1556
Encroach Node=12654
       1 1083.79  1366.5
Encroach Node=12594
       1 1083.79    1369
Encroach Node=12567
       1 1102.22  1381.5
Encroach Node=12547.34
       1 1128.31  1409.6
Encroach Node=12547.05
       1 1128.31  1409.6
Encroach Node=12488
       1 1110.23 1375.22
Encroach Node=12283
       1 1110.26 1375.22
Encroach Node=12225
       1 1009.75 1272.04
Encroach Node=12166
       1 1009.83 1271.98
Encroach Node=12152
       1  912.84 1181.01
Encroach Node=12124
       1  499.72  774.98
Encroach Node=12077
       1  414.47  683.72
Encroach Node=11941
       1  414.52  683.68
Encroach Node=11899
       1  722.48  979.83
Encroach Node=11695
       1 1257.49 1523.77
Encroach Node=11585
       1 1653.28 1921.43
Encroach Node=11377
       1    1877  2142.8
Encroach Node=10986
       1 2095.08  2372.5
Encroach Node=10917
       1 2263.02 2542.77
Encroach Node=10877
       1 2264.31  2544.7
Encroach Node=10649
       1 2080.09  2357.9
Encroach Node=10165
       1 2412.84  2689.3
Encroach Node=9751
       1 2059.45  2331.6
Encroach Node=9582
       1 1836.37  2113.7
Encroach Node=9532
       1 1787.24 2061.09
Encroach Node=9492
       1 1784.28 2060.97
Encroach Node=9442
       1 1773.95    2048
Encroach Node=9251
       1 1296.44  1568.1
Encroach Node=9082
       1 1715.66    1987
Encroach Node=8812
       1 1246.14  1522.7
Encroach Node=8638
       1 1055.97  1323.2
Encroach Node=8443
       1 1074.58  1322.4
Encroach Node=8301
       1  948.79 1389.86
Encroach Node=8210
       1   871.2 1502.22
Encroach Node=8168
       1  610.72  1293.5
Encroach Node=8155
       1  602.65    1278
Encroach Node=8130
       1  602.65 1277.42
Encroach Node=7766
       1  801.88 1421.38
Encroach Node=7168
       1 1078.13    1386
Encroach Node=6970
       1 1129.16    1440
Encroach Node=6769
       1 1091.54    1540
Encroach Node=6729
       1 1091.54 1506.74
Encroach Node=6623
       1  846.74 1326.35
Encroach Node=6456
       1  802.23 1277.84
Encroach Node=6414
       1  770.36 1326.88
Encroach Node=6396
       1  778.78  1335.3
Encroach Node=6296
       1  808.23  1429.5
Encroach Node=6248
       1  814.28 1461.94
Encroach Node=6149
       1  800.86 1314.58
Encroach Node=6064
       1  800.86 1314.58
Encroach Node=5901
       1  875.81  1391.6
Encroach Node=5776
       1  870.41 1328.01
Encroach Node=5599
       1  823.17 1203.42
Encroach Node=5399
       1  508.17     835
Encroach Node=5261
       1  380.48     695
Encroach Node=5014
       1  334.06     585
Encroach Node=4899
       1  338.33  529.36
Encroach Node=4689
       1  324.78     610
Encroach Node=4444
       1  328.78     630
Encroach Node=4331
       1  328.78     625
Encroach Node=4176
       1  244.45     603
Encroach Node=4027
       1  201.11     595
Encroach Node=3925
       1  191.25     580
Encroach Node=3612
       1  204.86     630
Encroach Node=3385
       1  213.56     670
Encroach Node=3093
       1     250     683
Encroach Node=2685
       1  271.99  658.03
Encroach Node=2552
       1  229.81  595.76
Encroach Node=2409
       1     260   510.2
Encroach Node=2192
       1  240.34  458.96
Encroach Node=1980
       1  184.95  408.33
Encroach Node=1763
       1  140.22  384.68
Encroach Node=1535
       1  136.68  353.44
Encroach Node=1394
       1  136.68  353.44
Encroach Node=1264
       1  139.37  362.78
Encroach Node=1032
       1  146.34  353.93
Encroach Node=808
       1   158.5  383.92
Encroach Node=667
       1  191.06  491.05
Encroach Node=500
       1     183     593
Encroach Node=472
       1     187     590
Encroach River=West Fork
Encroach Reach=wf4
Encroach Node=306141
       1    1424    2077
Encroach Node=304934
       1    1260    1665
Encroach Node=303800
       1 1291.01    1577
Encroach Node=303696
       1    1298  1580.9
Encroach Node=302918
       1    1170    1516
Encroach Node=301515
       1 1031.79    1805
Encroach Node=300650
       1 1029.91    1800
Encroach Node=299750
       1 1101.27    2000
Encroach Node=299057
       1 1118.42    1985
Encroach Node=299015
       1    1155    2025
Encroach Node=299009
       1    1180    2055
Encroach Node=298960
       1    1150    2035
Encroach Node=298126
       1    1122    1750
Encroach Node=297780
       1    1480    1850
Encroach Node=297741
       1    1495    1860
Encroach Node=297729
       1    1532    1885
Encroach Node=297678
       1    1532    1885
Encroach Node=297299
       1    1065    1309
Encroach Node=296731
       1 1100.69    1354
Encroach Node=296619
       1  1023.8 1267.32
Encroach Node=296581
       1 1024.02 1267.16
Encroach Node=296466
       1  1087.4    1319
Encroach Node=295601
       1  1084.1    1297
Encroach Node=294682
       1    1091    1297
Encroach Node=293700
       1    1085    1334
Encroach Node=293232
       1    1085    1317
Encroach Node=293128
       1 1028.49 1256.17
Encroach Node=293084
       1 1028.93 1255.93
Encroach Node=292982
       1    1089    1305
Encroach Node=292186
       1    1090 1301.21
Encroach Node=291311
       1    1090 1302.46
Encroach Node=290763
       1    1098    1295
Encroach Node=289753
       1    1098  1301.5
Encroach Node=288960
       1 1087.36    1306
Encroach Node=288923
       1 1087.45    1306
Encroach Node=288909
       1    1113    1313
Encroach Node=288865
       1    1123    1313
Encroach Node=288841
       1     242   458.2
Encroach Node=288673
       1   241.8   457.9
Encroach Node=288459
       1  314.94  543.41
Encroach Node=288273
       1  388.72  617.19
Encroach Node=287904
       1  424.65  659.64
Encroach Node=287531
       1  478.27  691.71
Encroach Node=287315
       1  893.81 1109.51
Encroach Node=287121
       1 1390.83 1603.57
Encroach Node=286943
       1 1418.93 1627.39
Encroach Node=286790
       1 1341.41 1554.28
Encroach Node=286597
       1 1091.26 1313.93
Encroach Node=286409
       1  1255.3    1470
Encroach Node=286264
       1   67.88     322
Encroach Node=286205
       1   83.24  288.83
Encroach Node=286013
       1   96.02   297.9
Encroach Node=285827
       1   94.05  300.61
Encroach Node=285640
       1   92.96  303.87
Encroach Node=285459
       1   91.94  303.04
Encroach Node=285240
       1   91.99  301.67
Encroach Node=284962
       1   89.07  294.48
Encroach Node=284710
       1    91.7  292.09
Encroach Node=284440
       1   84.21  296.37
Encroach Node=284120
       1   95.71  297.86
Encroach Node=283738
       1   97.51  299.85
Encroach Node=283362
       1   84.01  297.73
Encroach Node=283002
       1  283.79  509.18
Encroach Node=282728
       1  162.45   391.6
Encroach Node=282425
       1  158.36  380.16
Encroach Node=282100
       1  215.16  437.13
Encroach Node=281757
       1  258.97  477.63
Encroach Node=281586
       1     242  436.82
Encroach Node=281367
       1  107.34  414.64
Encroach Node=281317
       1  112.92  449.92
Encroach Node=281279
       1   66.14  352.56
Encroach Node=281259
       1   68.29  337.26
Encroach Node=281193
       1  162.71  406.63
Encroach Node=281069
       1  167.51  393.67
Encroach Node=280860
       1  158.53   359.4
Encroach Node=280594
       1  130.04  347.94
Encroach Node=280288
       1  257.47   475.8
Encroach Node=279978
       1  177.47  419.17
Encroach Node=279716
       1  138.71  377.93
Encroach Node=279530
       1  1088.6 1334.69
Encroach Node=279352
       1  777.23   999.9
Encroach Node=279021
       1  631.39  863.88
Encroach Node=278753
       1  576.93  843.87
Encroach Node=278512
       1  552.91  818.49
Encroach Node=278372
       1  406.12  681.29
Encroach Node=278273
       1  373.51  637.81
Encroach Node=278066
       1  361.58  627.81
Encroach Node=277882
       1  375.19  641.94
Encroach Node=277619
       1   399.4  662.63
Encroach Node=277257
       1  389.63  644.78
Encroach Node=276875
       1  374.28   637.8
Encroach Node=276534
       1  349.16  594.32
Encroach Node=276387
       1  312.32  520.47
Encroach Node=276324
       1  312.32  520.47
Encroach Node=276174
       1  198.41  438.93
Encroach Node=276064
       1  172.98  398.44
Encroach Node=275869
       1  145.27   359.9
Encroach Node=275742
       1  151.53  341.03
Encroach Node=275404
       1   153.5  348.34
Encroach Node=275021
       1  174.31  355.26
Encroach Node=274464
       1  186.99     425
Encroach Node=274320
       1  214.83     550
Encroach Node=274314
       1  214.83     550
Encroach Node=274273
       1  215.18     552
Encroach Node=274268
       1  215.18     552
Encroach Node=274089
       1  218.89     703
Encroach Node=273936
       1  227.19     675
Encroach Node=273635
       1  258.88  596.91
Encroach Node=273309
       1     295     596
Encroach Node=272958
       1     310     616
Encroach Node=272647
       1     300     625
Encroach Node=272324
       1     265     635
Encroach Node=272073
       1     260     630
Encroach Node=271755
       1     250     616
Encroach Node=271391
       1     248     620
Encroach Node=271022
       1     150     646
Encroach Node=270686
       1      89     674
Encroach Node=270374
       1   96.94    1032
Encroach Node=270065
       1    1480    2512
Encroach Node=269827
       1    1800    2885
Encroach Node=269732
       1  1453.6    2502
Encroach Node=269568
       1    1310    2352
Encroach Node=269272
       1    1125    2142
Encroach Node=269045
       1    1200    2186
Encroach Node=268631
       1    1275    2027
Encroach Node=268269
       1     950    1772
Encroach Node=267685
       1     750    1543
Encroach Node=267174
       1  724.39    1473
Encroach Node=266963
       1  686.35    1428
Encroach Node=266567
       1     750    1526
Encroach Node=266194
       1    1000    1927
Encroach Node=265554
       1    1200    2401
Encroach Node=264706
       1    1620    2996
Encroach Node=264149
       1    1730    2987
Encroach Node=263654
       1    1785    2991
Encroach Node=263416
       1    1670    2806
Encroach Node=262885
       1    1755    2679
Encroach Node=262637
       1    1565    2581
Encroach Node=262176
       1    1540    2535
Encroach Node=262091
       1    1523 2451.92
Encroach Node=261989
       1    1585 2451.89
Encroach Node=261964
       1    1510 2383.22
Encroach Node=261585
       1    1115    2020
Encroach Node=261188
       1    1025    1820
Encroach Node=260884
       1     925    1684
Encroach Node=260476
       1     795    1400
Encroach Node=260154
       1     685    1215
Encroach Node=259866
       1     555    1010
Encroach Node=259468
       1     345     700
Encroach Node=259059
       1      26   372.5
Encroach Node=258911
       1      26     358
Encroach Node=258689
       1     845 1116.55
Encroach Node=258409
       1  761.07 1091.58
Encroach Node=258186
       1  655.55 1038.93
Encroach Node=257970
       1  728.64 1164.78
Encroach Node=257763
       1     545 1002.58
Encroach Node=257540
       1     385  808.32
Encroach Node=257391
       1   251.1  647.46
Encroach Node=257177
       1  149.71   510.7
Encroach Node=257050
       1   122.7     557
Encroach Node=257008
       1     115     558
Encroach Node=256831
       1  132.58  512.64
Encroach Node=256674
       1  133.36  502.79
Encroach Node=256421
       1  131.96  470.56
Encroach Node=256161
       1  134.13  456.91
Encroach Node=255876
       1  140.35  447.75
Encroach Node=255668
       1  136.61  435.85
Encroach Node=255477
       1  138.49  416.04
Encroach Node=255240
       1   137.2  398.59
Encroach Node=255050
       1  128.86  362.27
Encroach Node=254923
       1  119.64   358.4
Encroach Node=254607
       1  155.07  588.65
Encroach Reach=wf3
Encroach Node=253939
       1   89.71     545
Encroach Node=253713
       1   77.78  387.44
Encroach Node=253684
       1   80.04     380
Encroach Node=253605
       1   76.69  327.73
Encroach Node=253517
       1   32.22  320.96
Encroach Node=253466
       1   33.22  324.77
Encroach Node=253311
       1   59.22  344.49
Encroach Node=253039
       1  107.39  390.45
Encroach Node=252896
       1  126.27  394.04
Encroach Node=252828
       1  136.15  417.02
Encroach Node=252702
       1     136  416.56
Encroach Node=252623
       1  146.48  442.21
Encroach Node=252522
       1  161.72   469.4
Encroach Node=252334
       1  194.51   497.8
Encroach Node=252164
       1  190.48  486.78
Encroach Node=251957
       1  186.25  494.99
Encroach Node=251646
       1  303.38   631.6
Encroach Node=251602
       1  324.92  655.33
Encroach Node=251552
       1  363.57  680.34
Encroach Node=251498
       1  388.12  698.91
Encroach Node=251478
       1   398.3  707.91
Encroach Node=251302
       1  431.95  719.29
Encroach Node=251168
       1  448.44  713.31
Encroach Node=251005
       1  420.31  692.95
Encroach Node=250795
       1  421.21  720.99
Encroach Node=250590
       1  379.84  689.47
Encroach Node=250304
       1  349.04   682.9
Encroach Node=250105
       1  330.52  645.88
Encroach Node=249860
       1  354.02   706.4
Encroach Node=249464
       1  389.73     703
Encroach Node=248969
       1  420.41     737
Encroach Node=248601
       1  408.82  715.25
Encroach Node=248281
       1  352.69     690
Encroach Node=247864
       1  265.82     596
Encroach Node=247550
       1     154  487.87
Encroach Node=247438
       1  151.11  480.12
Encroach Node=247071
       1  350.36  667.17
Encroach Node=246758
       1  453.48  824.65
Encroach Node=246657
       1  407.73     810
Encroach Node=246598
       1  376.72     794
Encroach Node=246486
       1  291.61     742
Encroach Node=246376
       1  207.68     689
Encroach Node=246135
       1  182.02     607
Encroach Node=245894
       1  111.58   502.8
Encroach Node=245570
       1   88.36  459.55
Encroach Node=245268
       1  132.32  461.81
Encroach Node=244971
       1  176.48  510.57
Encroach Node=244601
       1  144.84   482.7
Encroach Node=244320
       1  112.99  491.28
Encroach Node=244192
       1  107.65  457.68
Encroach Node=244046
       1  146.73  465.12
Encroach Node=243817
       1  142.54  466.25
Encroach Node=243538
       1  149.51  472.74
Encroach Node=243297
       1  172.41  509.01
Encroach Node=243005
       1  196.91  553.88
Encroach Node=242782
       1  219.26  591.14
Encroach Node=242570
       1  224.21  597.78
Encroach Node=242405
       1     221  586.86
Encroach Node=242152
       1     593 1012.99
Encroach Node=241937
       1  167.26  541.56
Encroach Node=241774
       1  174.38   499.6
Encroach Node=241724
       1  220.98  535.98
Encroach Node=241667
       1  142.81  474.65
Encroach Node=241637
       1  171.36  470.76
Encroach Node=241604
       1  171.36  470.76
Encroach Node=241564
       1  185.88  521.35
Encroach Node=241499
       1   56.49  396.46
Encroach Node=241485
       1   64.13     422
Encroach Node=241462
       1   64.13     422
Encroach Node=241447
       1   64.13  421.89
Encroach Node=241412
       1   36.49  376.83
Encroach Node=241386
       1    62.3  404.46
Encroach Node=241346
       1   63.34  401.52
Encroach Node=241328
       1   67.29  415.94
Encroach Node=241148
       1    1890    2370
Encroach Node=240938
       1    2740    3660
Encroach Node=240736
       1    2690    3720
Encroach Node=240563
       1    2760    3713
Encroach Node=240413
       1    2755    3710
Encroach Node=240247
       1    2510    3405
Encroach Node=240131
       1    2538    3306
Encroach Node=239943
       1 2583.24 3289.32
Encroach Node=239725
       1 2608.46 3231.22
Encroach Node=239391
       1 2397.03 2988.01
Encroach Node=239147
       1 2427.32 2934.89
Encroach Node=239002
       1 2418.02 2994.06
Encroach Node=238817
       1  2572.1 3067.16
Encroach Node=238734
       1 2618.16 2984.37
Encroach Node=238405
       1 2606.67 2969.95
Encroach Node=238109
       1 2508.03 2894.06
Encroach Node=238025
       1 2452.18 2750.91
Encroach Node=237781
       1  1557.2 1939.42
Encroach Node=237622
       1 1168.26 1552.75
Encroach Node=237406
       1  704.67 1074.43
Encroach Node=237005
       1  872.34 1263.64
Encroach Node=236685
       1  700.05 1179.18
Encroach Node=236323
       1  602.08 1172.34
Encroach Node=236074
       1  485.55 1089.03
Encroach Node=235625
       1  453.07  918.47
Encroach Node=235208
       1  398.37  870.61
Encroach Node=235058
       1  398.37  870.61
Encroach Node=235011
       1 1176.25 1717.28
Encroach Node=234833
       1  944.65 1501.56
Encroach Node=234605
       1   623.8 1113.01
Encroach Node=234374
       1   690.5 1124.61
Encroach Node=234112
       1  625.11 1101.14
Encroach Node=233766
       1  545.27 1100.94
Encroach Node=233474
       1  494.08 1019.24
Encroach Node=233258
       1  484.79 1005.11
Encroach Node=233029
       1  443.93  962.99
Encroach Node=232688
       1  451.62  909.06
Encroach Node=232559
       1  373.28  799.92
Encroach Node=232426
       1  419.31   820.8
Encroach Node=232296
       1  399.29  778.53
Encroach Node=232116
       1  394.12  754.45
Encroach Node=231974
       1  555.59  892.67
Encroach Node=231849
       1  726.03 1052.59
Encroach Node=231671
       1  896.14 1225.07
Encroach Node=231491
       1 1038.94 1387.24
Encroach Node=231299
       1  738.14 1076.12
Encroach Node=231219
       1  214.71  562.22
Encroach Node=231130
       1   97.24  618.94
Encroach Node=231049
       1   97.36     639
Encroach Node=230924
       1  175.17  764.47
Encroach Node=230880
       1  128.24     754
Encroach Node=230634
       1  128.24     754
Encroach Node=230574
       1   459.6  918.79
Encroach Node=230448
       1  413.31  873.01
Encroach Node=230199
       1  598.73 1057.79
Encroach Node=230042
       1  649.53 1081.14
Encroach Node=229933
       1  596.91 1013.21
Encroach Node=229746
       1  433.92  830.45
Encroach Node=229607
       1  562.39     937
Encroach Node=229455
       1  406.75  774.79
Encroach Node=229322
       1  252.57     719
Encroach Node=229237
       1  252.57     719
Encroach Node=229171
       1  496.11  930.26
Encroach Node=229064
       1  456.31  855.66
Encroach Node=229003
       1  468.33   844.9
Encroach Node=228848
       1  536.63  879.62
Encroach Node=228694
       1  635.75  989.55
Encroach Node=228544
       1  670.77 1023.84
Encroach Node=228303
       1  551.53  904.72
Encroach Node=227987
       1  421.21  780.93
Encroach Node=227941
       1   436.2  788.45
Encroach Node=227824
       1   884.6 1231.17
Encroach Node=227552
       1 1147.65 1641.46
Encroach Node=227034
       1 1559.74 2046.13
Encroach Node=226504
       1 2071.75  2551.3
Encroach Node=225979
       1 2324.42 2881.32
Encroach Node=225474
       1 2506.44 3132.02
Encroach Node=225215
       1 2520.53 3156.58
Encroach Node=224722
       1 2713.57 3316.61
Encroach Node=224241
       1 2883.27 3531.05
Encroach Node=223864
       1    2943    3615
Encroach Node=223686
       1 3009.42 3610.71
Encroach Node=223230
       1    2630  3231.2
Encroach Node=222936
       1    2020 3030.21
Encroach Node=222819
       1    1930 3064.43
Encroach Node=222768
       1    1878 3037.01
Encroach Node=222714
       1    1854    3120
Encroach Node=222506
       1    1810    3530
Encroach Node=222235
       1    1834    3674
Encroach Node=221540
       1    1780    3626
Encroach Node=221096
       1    1790    3706
Encroach Node=220847
       1    1958 3992.04
Encroach Node=220623
       1    1786    3870
Encroach Node=220360
       1    2019    4160
Encroach Node=220020
       1    2106    4230
Encroach Node=219656
       1    1690    3771
Encroach Node=219338
       1    1478    3470
Encroach Node=218953
       1    1750    3364
Encroach Node=218679
       1    1700    3312
Encroach Node=218595
       1    1739 3296.45
Encroach Node=218514
       1    1751  3439.3
Encroach Node=218485
       1    1718 3409.92
Encroach Node=218419
       1    1668 3409.71
Encroach Node=218372
       1    1673 3394.39
Encroach Node=218095
       1    1588 3744.83
Encroach Node=217842
       1    1312    3310
Encroach Node=217755
       1    1248    3275
Encroach Node=217585
       1    1240    3290
Encroach Node=217017
       1    1530    3730
Encroach Node=215964
       1    2000 4224.05
Encroach Node=215271
       1    2045 4591.66
Encroach Node=214805
       1 1631.81    4700
Encroach Node=213977
       1     790    4356
Encroach Node=212961
       1     960    4600
Encroach Node=212466
       1     870    4655
Encroach Node=211302
       1     900 5006.26
Encroach Node=210619
       1     990    5059
Encroach Node=210160
       1    1220    5345
Encroach Node=209857
       1    1470    5310
Encroach Node=209229
       1    1700    5175
Encroach Node=208743
       1    1810    5100
Encroach Node=208050
       1    1846    5136
Encroach Node=206389
       1    1910    4992
Encroach Node=206158
       1    1710 4914.25
Flow Ratio Tolerance=0.1
Flow Ratio Min Ratio=0.5
Flow Ratio Max Ratio=4
Flow Ratio Max Iterations= 10
BEGIN DESCRIPTION:
Existing Model
This plan is valid upstream of West Fork cross-section 206218 for the West Fork, Elm Fork, and Trinity River Main Stem.  This plan represents the FEMA Floodway using the 1% AEP peak flows and the NFIP 10%, 4%, 2%, 1%, 1%+ geometry.
END DESCRIPTION:
Computation Interval=1HOUR
Output Interval=1HOUR
Instantaneous Interval=1HOUR
Mapping Interval=1HOUR
Computation Time Step Use Courant=        0
Computation Time Step Use Time Series=    0
Computation Time Step Count To Double=0
Computation Time Step Max Doubling=0
Computation Time Step Max Halving=0
Computation Time Step Residence Courant=0
Run HTab= 0
Run UNet= 0
Run Sediment= 0
Run PostProcess= 0
Run WQNet= 0
Run RASMapper= 0
UNET Theta= 1
UNET Theta Warmup= 1
UNET ZTol= 0.02
UNET ZSATol= 0.05
UNET MxIter= 20
UNET Max Iter WO Improvement= 0
UNET MaxInSteps= 0
UNET DtIC= 0
UNET DtMin= 0
UNET MaxCRTS= 20
UNET WFStab= 2
UNET SFStab= 1
UNET WFX= 1
UNET SFX= 1
UNET Gravity=32.17405
UNET 1D Methodology=Finite Difference
UNET DSS MLevel= 4
UNET Pardiso=0
UNET DZMax Abort= 100
UNET Use Existing IB Tables=-1
UNET Froude Reduction=False
UNET Froude Limit= 1
UNET Froude Power= 10
UNET D1 Cores= 0
UNET WindReference=Eulerian
UNET WindDragFormulation=Hsu (1988)
UNET D2 Coriolis=0
UNET D2 Cores= 0
UNET D2 Theta= 1
UNET D2 Theta Warmup= 1
UNET D2 Z Tol= 0.01
UNET D2 Volume Tol= 0.01
UNET D2 Max Iterations= 20
UNET D2 Advanced Convergence=0
UNET D2 WS Max Tol=0.15
UNET D2 WS RMS Tol=0.002
UNET D2 WS Stall Tol=1
UNET D2 Equation= 0
UNET D2 RampUpFraction=0.1
UNET D2 TimeSlices= 1
UNET D2 Turbulence Formulation=Non-Conservative (original)
UNET D2 Eddy Viscosity=0.3
UNET D2 Transverse Eddy Viscosity=0.3
UNET D2 Smagorinsky Mixing=0
UNET D2 BCVolumeCheck=0
UNET D2 Cores=0
UNET D2 SolverType=PARDISO (Direct)
UNET D2 Minimum Iterations= 3
UNET D2 Maximum Iterations= 30
UNET D2 Restart Number= 10
UNET D2 Relaxation Coeff=1.3
UNET D2 SOR Precondition Iterations= 10
UNET D2 ILUT Maximum Fill= 8
UNET D2 ILUT Tolerance=1E-08
UNET D2 Convergence Tolerance=0.00001
PS Theta= 1
PS WS Tol= 0.01
PS Volume Tol= 0.01
PS Max Iterations= 20
PS Equation= 0
PS Advance Time Step=-1
PS Target Courant=0.9
PS Time Slices= 1
PS Iterate With 2D=0
PS Project Initial WSE from DS=-1
PS Ramp Up Initial WSE from US=-1
PS Cores=0
UNET D1D2 MaxIter= 0
UNET D1D2 ZTol=0.01
UNET D1D2 QTol=0.1
UNET D1D2 MinQTol=1
Write IC File= 0
Write IC File at Fixed DateTime=0
Write IC File at Sim End=0
Echo Input=False
Echo Parameters=False
Echo Output=False
Write Detailed= 0
HDF Write Warmup=0
HDF Write Time Slices=0
HDF Flush=0
HDF Compression= 1
HDF Chunk Size= 1
HDF Spatial Parts= 1
HDF Use Max Rows=0
HDF Fixed Rows= 1
Calibration Method= 0
Calibration Iterations= 20
Calibration Max Change=0.05
Calibration Tolerance=0.2
Calibration Maximum=1.5
Calibration Minimum=0.5
Calibration Optimization Method= 1
WQ AD Non Conservative
WQ ULTIMATE=-1
WQ Max Comp Step=1HOUR
WQ Output Interval=15MIN
WQ Output Selected Increments= 0
WQ Create Restart=0
WQ Fixed Restart=0
WQ System Summary=0
WQ Write To DSS=0
Sorting and Armoring Iterations= 10
XS Update Threshold= 0.02
Bed Roughness Predictor= 0
Processes Affected by Predictor=Sediment Only
Hydraulics Update Threshold= 0.02
Energy Slope Method= 2
Volume Change Method= 0
Sediment Retention Method= 0
Sediment TS Multiplier= 1
Warm Up Method= 0
XS Weighting Method= 0
Number of US Weighted Cross Sections= 1
Number of DS Weighted Cross Sections= 1
Upstream XS Weight=0.25
Main XS Weight=0.5
Downstream XS Weight=0.25
Number of DS XS's Weighted with US Boundary= 1
Upstream Boundary Weight= 1
Weight of XSs Associated with US Boundary= 0
Number of US XS's Weighted with DS Boundary= 1
Downstream Boundary Weight= 0.5
Weight of XSs Associated with DS Boundary= 0.5
Percentile Method= 0
Sediment Output Level= 4
Mass or Volume Output= 0
Output Increment Type= 1
Profile and TS Output Increment= 10
Transport Output Increment 1
XS Output Flag= 0
XS Output Increment= 10
Read HDF5 Sediment Hotstart= 0
Sediment Hotstart Type= 0
Write Gradation File= 0
Read Gradation Hotstart= 0
Write HDF5 File= 1
Write Binary Output= 1
Write DSS Sediment File= 0
DSS Sediment Output Type= 1
SV Curve= 0
Specific Gage Flag= 0
Subcell Erosion Methods= 0
Subcell Deposition Methods= 0
Advection Scheme= 1
Matrix Solver= 0
Implicit Weighting Factor= 1
Maximum Outer Loop Convergence Iterations= 5
Convergence Maximum Absolute= 0.001
Convergence RMSE= 0.0001
Grain Fractions Max Abs Error= 0.001
Max Subgrid Regions= 1
Max Subgrid Length Scale= 3.402823E+38
Initial Layer Thickness= 3
Min Layer Thickness= 0.1
Max Layer Thickness= 6
Number of Layers= 5

--- CDC_Consolidated_Model.p06 (plan) ---

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Plan Title=Exist: 1%+ AEP [WF/EF/TRMS]
Program Version=6.60
Short Identifier=Existing Plan 6
Geom File=g04
Flow File=f06
Flow Ratio Tolerance=0.1
Flow Ratio Min Ratio=0.5
Flow Ratio Max Ratio=4
Flow Ratio Max Iterations= 10
Existing Model
This plan is valid downstream of West Fork cross-section 206218 for the West Fork, Elm Fork, and Trinity River Main Stem.  This plan represents the 1%+ AEP peak flows and geometry.
UNET Gravity=32.17405
UNET WindReference=Eulerian
UNET WindDragFormulation=Hsu (1988)
UNET D2 Advanced Convergence=0
UNET D2 WS Max Tol=0.15
UNET D2 WS RMS Tol=0.002
UNET D2 WS Stall Tol=1
UNET D2 Turbulence Formulation=Non-Conservative (original)
UNET D2 Eddy Viscosity=0.3
UNET D2 Transverse Eddy Viscosity=0.3
UNET D2 Smagorinsky Mixing=0
UNET D2 Cores=0
UNET D2 SolverType=PARDISO (Direct)
UNET D2 Minimum Iterations= 3
UNET D2 Maximum Iterations= 30
UNET D2 Restart Number= 10
UNET D2 Relaxation Coeff=1.3
UNET D2 SOR Precondition Iterations= 10
UNET D2 ILUT Maximum Fill= 8
UNET D2 ILUT Tolerance=1E-08
UNET D2 Convergence Tolerance=0.00001
PS Theta= 1
PS WS Tol= 0.01
PS Volume Tol= 0.01
PS Max Iterations= 20
PS Equation= 0
PS Advance Time Step=-1
PS Target Courant=0.9
PS Time Slices= 1
PS Iterate With 2D=0
PS Project Initial WSE from DS=-1
PS Ramp Up Initial WSE from US=-1
PS Cores=0
DSS File=dss
Processes Affected by Predictor=Sediment Only
Energy Slope Method= 2
Sediment TS Multiplier= 1
Warm Up Method= 0
Transport Output Increment 1
Read HDF5 Sediment Hotstart= 0
Sediment Hotstart Type= 0
DSS Sediment Output Type= 1
Subcell Erosion Methods= 0
Subcell Deposition Methods= 0
Advection Scheme= 1
Matrix Solver= 0
Implicit Weighting Factor= 1
Maximum Outer Loop Convergence Iterations= 5
Convergence Maximum Absolute= 0.001
Convergence RMSE= 0.0001
Grain Fractions Max Abs Error= 0.001
Max Subgrid Regions= 1
Max Subgrid Length Scale= 3.402823E+38
Initial Layer Thickness= 3
Min Layer Thickness= 0.1
Max Layer Thickness= 6
Number of Layers= 5

--- CDC_Consolidated_Model.p12 (plan) ---

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Plan Title=CDC: 50% to 1% AEP [WF/EF/TRMS]
Short Identifier=CDC Plan 12
Geom File=g12
Flow File=f12
Secant Critical Depth
This plan is valid downstream of West Fork cross-section 206218 for the West Fork, Elm Fork, and Trinity River Main Stem.  This plan represents the 50%, 20%, 10%, 4%, 2%, 1% AEP peak flows and geometry.
DSS File=dss

--- CDC_Consolidated_Model.p13 (plan) ---

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Plan Title=CDC: 0.2% AEP, SPF [WF/EF/TRMS]
Short Identifier=CDC Plan 13
Geom File=g13
Flow File=f13
This plan is valid downstream of West Fork cross-section 206218 for the West Fork, Elm Fork, and Trinity River Main Stem.  This plan represents the 0.2% AEP and SPF peak flows and geometry.
DSS File=dss

--- CDC_Consolidated_Model.f11 (steady flow) ---

Flow Title=CDC: 50% to 0.2% AEP, SPF [WF/CF]
Program Version=6.10
BEGIN FILE DESCRIPTION:
CDC: 50%, 20%, 10%, 4%, 2%, 1%, 0.2% ACE (Annual Exceedance Probability) and SPF peak flows
END FILE DESCRIPTION:
Number of Profiles= 8
Profile Names=50% AEP,20% AEP,10% AEP,4% AEP,2% AEP,1% AEP,0.2% AEP,SPF
River Rch & RM=Clear Fork,cf              ,65437
       1       1       1       1       1       1       1       1
River Rch & RM=Clear Fork,cf              ,60344
    3100    4700    6200    8200    9800   13000   46000   72000
River Rch & RM=Clear Fork,cf              ,40990
   13500   20000   26500   34500   41500   48500   61500   95500
River Rch & RM=Clear Fork,cf              ,35052
   13500   20500   27000   35000   42500   50000   66500   94500
River Rch & RM=Clear Fork,cf              ,8335
   13500   20500   26500   34000   41000   48500   66000   93000
River Rch & RM=West Fork,wf4             ,305599.5
    8100   13500   15000   23500   29000   35000   54000   56500
River Rch & RM=West Fork,wf4             ,289624.5
    8200   13500   15000   23500   28500   35000   54000   63500
River Rch & RM=West Fork,wf3             ,253818.1
   17000   25500   34500   48000   59000   69500  107000  136000
River Rch & RM=West Fork,wf3             ,248160.
   17000   25500   35000   48000   59000   69000  107000  136000
River Rch & RM=West Fork,wf3             ,241815.4
   18000   27000   36000   49500   60500   71500  111000  140000
River Rch & RM=West Fork,wf3             ,234252.7
   17500   28000   37000   49500   59500   68000  112000  143000
River Rch & RM=West Fork,wf3             ,221418.5
   21000   35500   48000   43500   74500   83500  133000  165000
River Rch & RM=West Fork,wf3             ,207998.0
   16500   28500   39500   55000   67000   78000  123000  154000
Boundary for River Rch & Prof#=Clear Fork,cf              , 1
Up Type= 0
Dn Type= 0
Boundary for River Rch & Prof#=Clear Fork,cf              , 2
Up Type= 0
Dn Type= 0
Boundary for River Rch & Prof#=Clear Fork,cf              , 3
Up Type= 0
Dn Type= 0
Boundary for River Rch & Prof#=Clear Fork,cf              , 4
Up Type= 0
Dn Type= 0
Boundary for River Rch & Prof#=Clear Fork,cf              , 5
Up Type= 0
Dn Type= 0
Boundary for River Rch & Prof#=Clear Fork,cf              , 6
Up Type= 0
Dn Type= 0
Boundary for River Rch & Prof#=Clear Fork,cf              , 7
Up Type= 0
Dn Type= 0
Boundary for River Rch & Prof#=Clear Fork,cf              , 8
Up Type= 0
Dn Type= 0
Boundary for River Rch & Prof#=West Fork,wf4             , 1
Up Type= 0
Dn Type= 0
Boundary for River Rch & Prof#=West Fork,wf4             , 2
Up Type= 0
Dn Type= 0
Boundary for River Rch & Prof#=West Fork,wf4             , 3
Up Type= 0
Dn Type= 0
Boundary for River Rch & Prof#=West Fork,wf4             , 4
Up Type= 0
Dn Type= 0
Boundary for River Rch & Prof#=West Fork,wf4             , 5
Up Type= 0
Dn Type= 0
Boundary for River Rch & Prof#=West Fork,wf4             , 6
Up Type= 0
Dn Type= 0
Boundary for River Rch & Prof#=West Fork,wf4             , 7
Up Type= 0
Dn Type= 0
Boundary for River Rch & Prof#=West Fork,wf4             , 8
Up Type= 0
Dn Type= 0
Boundary for River Rch & Prof#=West Fork,wf3             , 1
Up Type= 0
Dn Type= 4
Dn Rating Curve # Pts= 10
       0     472   16500  501.18   28500  506.15   39500  507.52   55000  510.08
   67000  511.62   78000  512.88  123000  517.23  154000  519.78  180000   521.5
Boundary for River Rch & Prof#=West Fork,wf3             , 2
Up Type= 0
Dn Type= 4
Boundary for River Rch & Prof#=West Fork,wf3             , 3
Up Type= 0
Dn Type= 4
Boundary for River Rch & Prof#=West Fork,wf3             , 4
Up Type= 0
Dn Type= 4
Boundary for River Rch & Prof#=West Fork,wf3             , 5
Up Type= 0
Dn Type= 4
Boundary for River Rch & Prof#=West Fork,wf3             , 6
Up Type= 0
Dn Type= 4
Boundary for River Rch & Prof#=West Fork,wf3             , 7
Up Type= 0
Dn Type= 4
Boundary for River Rch & Prof#=West Fork,wf3             , 8
Up Type= 0
Dn Type= 4
Set Internal Change=Clear Fork      ,cf              ,43262   , 6 , 3 ,611.2
Observed RC=Fort Worth Gage,West Fork       ,wf3             ,251524.5,0
Observed RC Desc=Data from USGS June 2007
Observed RC Data= 14
  519.54       0     520      24     521     923     522    2710     523    5550
     524    9310     525   13600     526   18400     527   23500     528   29100
     529   35200   529.1   35900   529.2   36500  529.24   36800
Observed RC Point Data= 0
Observed RC=Clear Fork Gage,Clear Fork      ,cf              ,12901.55,0
Observed RC Desc=Data from USGS June 2007
Observed RC Data= 24
  540.97       0     541     .06   541.5      23     542     207   542.5     767
     543    1350   543.5    2080     544    3030   544.5    4150     545    5430
   545.5    6850     546    8310   546.5    9800     547   11400   547.5   13000
     548   14700   548.5   16400     549   18200   549.5   20100   549.6   20500
   549.7   20900   549.8   21300   549.9   21700  549.91   21700
Observed RC Point Data= 0
DSS Import GetInterval= 0
DSS Import GetPeak= 0
DSS Import FillOption= 0
