HEC-RAS study CDC_Consolidated_Model.prj: Upper Trinity CDC Consolidated Model

--- CDC_Consolidated_Model.f01 (steady flow) ---

Flow Title=Exist: 10%, 4%, 2%, 1% AEP [WF/EF/TRMS]
Program Version=6.60
BEGIN FILE DESCRIPTION:
Existing: 10%, 4%, 2%, 1% AEP (Annual Exceedance Probability) peak flows
END FILE DESCRIPTION:
Number of Profiles= 4
Profile Names=10% AEP,4% AEP,2% AEP,1% AEP
River Rch & RM=Elm Fork,ef6             ,153340
    7000    7000    7000    7000
River Rch & RM=Elm Fork,ef5             ,147501
    7000    7000   10200   21000
River Rch & RM=Elm Fork,ef4             ,138526
    3500    3500    4500    7000
River Rch & RM=Elm Fork,ef3             ,125671
    7000    7000   10200   21000
River Rch & RM=Elm Fork,ef3             ,118745
    8016   10132   12123   21000
River Rch & RM=Elm Fork,ef3             ,112469
    8126   10304   12372   21000
River Rch & RM=Elm Fork,ef3             ,107977
   23148   30680   36841   44597
River Rch & RM=Elm Fork,ef3             ,102709
   21555   28547   34831   43553
River Rch & RM=Elm Fork,ef3             ,93155
   20886   27657   33357   41276
River Rch & RM=Elm Fork,ef3             ,80596
   21694   29314   35266   43419
River Rch & RM=Elm Fork,ef3             ,64635
   20918   28582   34935   42825
River Rch & RM=Elm Fork,ef3             ,53311
   20918   28582   34935   42825
River Rch & RM=Elm Fork,ef2             ,48931
   1940025639.9129869.43   32000
River Rch & RM=Elm Fork,ef1             ,31628
   20918   28582   34935   42825
River Rch & RM=Elm Fork,ef1             ,30779
   19368   26437   33321   41462
River Rch & RM=Elm Fork,ef1             ,24559
   18991   25902   32912   41153
River Rch & RM=Elm Fork,ef1             ,17640
   18808   25541   32587   41366
River Rch & RM=Elm Fork L-Spill,efl             ,15577
       1    3300   10200   21000
River Rch & RM=Elm Fork Split1,efs1            ,9111
 1517.752942.2845065.57710824.85
River Rch & RM=Elm Fork Split2,efs2            ,133117
    3500    3500    6700   14000
River Rch & RM=Main Stem,ms              ,148139
   44240   71609   95040  118755
River Rch & RM=Main Stem,ms              ,110079
   39824   66882   88450  113234
River Rch & RM=Main Stem,ms              ,82348
   46951   70459   93071  118845
River Rch & RM=Main Stem,ms              ,76808
   45821   69577   91872  117706
River Rch & RM=Main Stem,ms              ,53576
   45821   69577   91872  117706
River Rch & RM=Main Stem,ms              ,51043
   45821   69577   91872  117706
River Rch & RM=West Fork,wf3             ,206158
   30115   45468   57609   68794
River Rch & RM=West Fork,wf3             ,184441
   36962   58148   72202   86097
River Rch & RM=West Fork,wf3             ,162387
   33584   53735   67624   82295
River Rch & RM=West Fork,wf3             ,140843
   40061   62254   78697   97693
River Rch & RM=West Fork,wf3             ,133374
   38091   59674   75804   95167
River Rch & RM=West Fork,wf3             ,123707
   38431   60455   76857   96559
River Rch & RM=West Fork,wf3             ,116017
   37408   59515   75891   95854
River Rch & RM=West Fork,wf3f            ,112687
    4808   19000   30891   47926
River Rch & RM=West Fork,wf3e            ,111697
   32600   40515   45000   47928
River Rch & RM=West Fork,wf3d            ,107732
   37408   59515   75891   95854
River Rch & RM=West Fork,wf3d            ,96217
   36153   57871   73945   93111
River Rch & RM=West Fork,wf3b            ,84526
   20607   30440   38895   49000
River Rch & RM=West Fork,wf3c            ,80116
   15546   27431   35050   44111
River Rch & RM=West Fork,wf3a            ,74827
   36153   57871   73945   93111
River Rch & RM=West Fork,wf2             ,53716
   36103   56871   70445   86111
River Rch & RM=West Fork,wf2             ,35195
   34865   55867   69039   84997
River Rch & RM=West Fork,wf1             ,34256
   34915   56867   72539   91997
River Rch & RM=West Fork,wf1             ,24876
   37215   61585   78568   95062
River Rch & RM=West Fork,wf1             ,11909
   32384   57555   74991   94443
River Rch & RM=West Fork,wf1             ,1494
   31656   56151   73823   93993
River Rch & RM=West Fork Split,wfs             ,56034
      50    1000    3500    7000
Boundary for River Rch & Prof#=Elm Fork,ef6             , 1
Up Type= 3
Up Slope=0.001
Dn Type= 0
Boundary for River Rch & Prof#=Elm Fork,ef6             , 2
Up Type= 3
Up Slope=0.001
Dn Type= 0
Boundary for River Rch & Prof#=Elm Fork,ef6             , 3
Up Type= 3
Up Slope=0.001
Dn Type= 0
Boundary for River Rch & Prof#=Elm Fork,ef6             , 4
Up Type= 3
Up Slope=0.001
Dn Type= 0
Boundary for River Rch & Prof#=Elm Fork,ef5             , 1
Up Type= 0
Dn Type= 0
Boundary for River Rch & Prof#=Elm Fork,ef5             , 2
Up Type= 0
Dn Type= 0
Boundary for River Rch & Prof#=Elm Fork,ef5             , 3
Up Type= 0
Dn Type= 0
Boundary for River Rch & Prof#=Elm Fork,ef5             , 4
Up Type= 0
Dn Type= 0
Boundary for River Rch & Prof#=Elm Fork,ef4             , 1
Up Type= 0
Dn Type= 0
Boundary for River Rch & Prof#=Elm Fork,ef4             , 2
Up Type= 0
Dn Type= 0
Boundary for River Rch & Prof#=Elm Fork,ef4             , 3
Up Type= 0
Dn Type= 0
Boundary for River Rch & Prof#=Elm Fork,ef4             , 4
Up Type= 0
Dn Type= 0
Boundary for River Rch & Prof#=Elm Fork,ef3             , 1
Up Type= 0
Dn Type= 0
Boundary for River Rch & Prof#=Elm Fork,ef3             , 2
Up Type= 0
Dn Type= 0
Boundary for River Rch & Prof#=Elm Fork,ef3             , 3
Up Type= 0
Dn Type= 0
Boundary for River Rch & Prof#=Elm Fork,ef3             , 4
Up Type= 0
Dn Type= 0
Boundary for River Rch & Prof#=Elm Fork,ef2             , 1
Up Type= 0
Dn Type= 0
Boundary for River Rch & Prof#=Elm Fork,ef2             , 2
Up Type= 0
Dn Type= 0
Boundary for River Rch & Prof#=Elm Fork,ef2             , 3
Up Type= 0
Dn Type= 0
Boundary for River Rch & Prof#=Elm Fork,ef2             , 4
Up Type= 0
Dn Type= 0
Boundary for River Rch & Prof#=Elm Fork,ef1             , 1
Up Type= 0
Dn Type= 1
Dn Known WS=415.12
Boundary for River Rch & Prof#=Elm Fork,ef1             , 2
Up Type= 0
Dn Type= 1
Dn Known WS=418.34
Boundary for River Rch & Prof#=Elm Fork,ef1             , 3
Up Type= 0
Dn Type= 1
Dn Known WS=420.73
Boundary for River Rch & Prof#=Elm Fork,ef1             , 4
Up Type= 0
Dn Type= 1
Dn Known WS=422.97
Boundary for River Rch & Prof#=Elm Fork L-Spill,efl             , 1
Up Type= 3
Up Slope=0.0022
Dn Type= 0
Boundary for River Rch & Prof#=Elm Fork L-Spill,efl             , 2
Up Type= 3
Up Slope=0.0022
Dn Type= 0
Boundary for River Rch & Prof#=Elm Fork L-Spill,efl             , 3
Up Type= 3
Up Slope=0.0022
Dn Type= 0
Boundary for River Rch & Prof#=Elm Fork L-Spill,efl             , 4
Up Type= 3
Up Slope=0.0022
Dn Type= 0
Boundary for River Rch & Prof#=Elm Fork Split1,efs1            , 1
Up Type= 0
Dn Type= 0
Boundary for River Rch & Prof#=Elm Fork Split1,efs1            , 2
Up Type= 0
Dn Type= 0
Boundary for River Rch & Prof#=Elm Fork Split1,efs1            , 3
Up Type= 0
Dn Type= 0
Boundary for River Rch & Prof#=Elm Fork Split1,efs1            , 4
Up Type= 0
Dn Type= 0
Boundary for River Rch & Prof#=Elm Fork Split2,efs2            , 1
Up Type= 0
Dn Type= 0
Boundary for River Rch & Prof#=Elm Fork Split2,efs2            , 2
Up Type= 0
Dn Type= 0
Boundary for River Rch & Prof#=Elm Fork Split2,efs2            , 3
Up Type= 0
Dn Type= 0
Boundary for River Rch & Prof#=Elm Fork Split2,efs2            , 4
Up Type= 0
Dn Type= 0
Boundary for River Rch & Prof#=Main Stem,ms              , 1
Up Type= 0
Dn Type= 1
Dn Known WS=385.8
Boundary for River Rch & Prof#=Main Stem,ms              , 2
Up Type= 0
Dn Type= 1
Dn Known WS=389.99
Boundary for River Rch & Prof#=Main Stem,ms              , 3
Up Type= 0
Dn Type= 1
Dn Known WS=392.38
Boundary for River Rch & Prof#=Main Stem,ms              , 4
Up Type= 0
Dn Type= 1
Dn Known WS=394.69
Boundary for River Rch & Prof#=West Fork,wf3             , 1
Up Type= 0
Dn Type= 0
Boundary for River Rch & Prof#=West Fork,wf3             , 2
Up Type= 0
Dn Type= 0
Boundary for River Rch & Prof#=West Fork,wf3             , 3
Up Type= 0
Dn Type= 0
Boundary for River Rch & Prof#=West Fork,wf3             , 4
Up Type= 0
Dn Type= 0
Boundary for River Rch & Prof#=West Fork,wf3f            , 1
Up Type= 0
Dn Type= 0
Boundary for River Rch & Prof#=West Fork,wf3f            , 2
Up Type= 0
Dn Type= 0
Boundary for River Rch & Prof#=West Fork,wf3f            , 3
Up Type= 0
Dn Type= 0
Boundary for River Rch & Prof#=West Fork,wf3f            , 4
Up Type= 0
Dn Type= 0
Boundary for River Rch & Prof#=West Fork,wf3e            , 1
Up Type= 0
Dn Type= 0
Boundary for River Rch & Prof#=West Fork,wf3e            , 2
Up Type= 0
Dn Type= 0
Boundary for River Rch & Prof#=West Fork,wf3e            , 3
Up Type= 0
Dn Type= 0
Boundary for River Rch & Prof#=West Fork,wf3e            , 4
Up Type= 0
Dn Type= 0
Boundary for River Rch & Prof#=West Fork,wf3d            , 1
Up Type= 0
Dn Type= 0
Boundary for River Rch & Prof#=West Fork,wf3d            , 2
Up Type= 0
Dn Type= 0
Boundary for River Rch & Prof#=West Fork,wf3d            , 3
Up Type= 0
Dn Type= 0
Boundary for River Rch & Prof#=West Fork,wf3d            , 4
Up Type= 0
Dn Type= 0
Boundary for River Rch & Prof#=West Fork,wf3b            , 1
Up Type= 0
Dn Type= 0
Boundary for River Rch & Prof#=West Fork,wf3b            , 2
Up Type= 0
Dn Type= 0
Boundary for River Rch & Prof#=West Fork,wf3b            , 3
Up Type= 0
Dn Type= 0
Boundary for River Rch & Prof#=West Fork,wf3b            , 4
Up Type= 0
Dn Type= 0
Boundary for River Rch & Prof#=West Fork,wf3c            , 1
Up Type= 0
Dn Type= 0
Boundary for River Rch & Prof#=West Fork,wf3c            , 2
Up Type= 0
Dn Type= 0
Boundary for River Rch & Prof#=West Fork,wf3c            , 3
Up Type= 0
Dn Type= 0
Boundary for River Rch & Prof#=West Fork,wf3c            , 4
Up Type= 0
Dn Type= 0
Boundary for River Rch & Prof#=West Fork,wf3a            , 1
Up Type= 0
Dn Type= 0
Boundary for River Rch & Prof#=West Fork,wf3a            , 2
Up Type= 0
Dn Type= 0
Boundary for River Rch & Prof#=West Fork,wf3a            , 3
Up Type= 0
Dn Type= 0
Boundary for River Rch & Prof#=West Fork,wf3a            , 4
Up Type= 0
Dn Type= 0
Boundary for River Rch & Prof#=West Fork,wf2             , 1
Up Type= 0
Dn Type= 0
Boundary for River Rch & Prof#=West Fork,wf2             , 2
Up Type= 0
Dn Type= 0
Boundary for River Rch & Prof#=West Fork,wf2             , 3
Up Type= 0
Dn Type= 0
Boundary for River Rch & Prof#=West Fork,wf2             , 4
Up Type= 0
Dn Type= 0
Boundary for River Rch & Prof#=West Fork,wf1             , 1
Up Type= 0
Dn Type= 0
Boundary for River Rch & Prof#=West Fork,wf1             , 2
Up Type= 0
Dn Type= 0
Boundary for River Rch & Prof#=West Fork,wf1             , 3
Up Type= 0
Dn Type= 0
Boundary for River Rch & Prof#=West Fork,wf1             , 4
Up Type= 0
Dn Type= 0
Boundary for River Rch & Prof#=West Fork Split,wfs             , 1
Up Type= 0
Dn Type= 0
Boundary for River Rch & Prof#=West Fork Split,wfs             , 2
Up Type= 0
Dn Type= 0
Boundary for River Rch & Prof#=West Fork Split,wfs             , 3
Up Type= 0
Dn Type= 0
Boundary for River Rch & Prof#=West Fork Split,wfs             , 4
Up Type= 0
Dn Type= 0
DSS Import GetInterval= 0
DSS Import GetPeak= 0
DSS Import FillOption= 0

--- CDC_Consolidated_Model.f02 (steady flow) ---

Flow Title=Exist: 0.2% AEP [WF/EF/TRMS]
Program Version=6.60
BEGIN FILE DESCRIPTION:
Existing: 0.2% ACE (Annual Exceedance Probability) peak flows
END FILE DESCRIPTION:
Number of Profiles= 1
Profile Names=0.2% AEP
River Rch & RM=Elm Fork,ef6             ,153340
    7000
River Rch & RM=Elm Fork,ef5             ,147501
   57000
River Rch & RM=Elm Fork,ef4             ,138526
    9500
River Rch & RM=Elm Fork,ef3             ,125671
   57000
River Rch & RM=Elm Fork,ef3             ,118745
   57000
River Rch & RM=Elm Fork,ef3             ,112469
   57000
River Rch & RM=Elm Fork,ef3             ,107977
   65779
River Rch & RM=Elm Fork,ef3             ,102709
   65779
River Rch & RM=Elm Fork,PGBT split west ,97191
   50000
River Rch & RM=Elm Fork,PGBT split east ,98000
15778.59
River Rch & RM=Elm Fork,ef3 ds          ,87661
   65779
River Rch & RM=Elm Fork,ef3 ds          ,87553
   61763
River Rch & RM=Elm Fork,ef3 ds          ,80596
   64587
River Rch & RM=Elm Fork,ef3 ds          ,72731
   64587
River Rch & RM=Elm Fork,ef3 ds          ,53311
   61427
River Rch & RM=Elm Fork,ef3 ds          ,48931
   61427
River Rch & RM=Elm Fork,ef3 ds          ,31628
   59479
River Rch & RM=Elm Fork,ef3 ds          ,23599
   59223
River Rch & RM=Elm Fork,ef3 ds          ,18646
   59223
River Rch & RM=Elm Fork L-Spill,efl             ,15577
   57000
River Rch & RM=Elm Fork Split2,efs2            ,133117
   47500
River Rch & RM=Main Stem,ms              ,148139
  190361
River Rch & RM=Main Stem,ms              ,110079
  182028
River Rch & RM=Main Stem,ms              ,82348
  191122
River Rch & RM=Main Stem,ms              ,76808
  189516
River Rch & RM=Main Stem,ms              ,53576
  189516
River Rch & RM=Main Stem,ms              ,51043
  189516
River Rch & RM=West Fork,wf              ,206158
  110745
River Rch & RM=West Fork,wf              ,184441
  132878
River Rch & RM=West Fork,wf              ,162387
  128817
River Rch & RM=West Fork,wf              ,140843
  158664
River Rch & RM=West Fork,wf              ,133374
  155546
River Rch & RM=West Fork,wf              ,123707
  158034
River Rch & RM=West Fork,wf              ,116017
  156592
River Rch & RM=West Fork,wf              ,107732
  156592
River Rch & RM=West Fork,wf              ,96217
  153715
River Rch & RM=West Fork,wf              ,74827
  153715
River Rch & RM=West Fork,wf              ,53716
  153715
River Rch & RM=West Fork,wf              ,35195
  150839
River Rch & RM=West Fork,wf              ,34256
  150839
River Rch & RM=West Fork,wf              ,24876
  161582
River Rch & RM=West Fork,wf              ,11909
  153340
River Rch & RM=West Fork,wf              ,1494
  152393
Boundary for River Rch & Prof#=Elm Fork,ef6             , 1
Up Type= 3
Up Slope=0.001
Dn Type= 0
Boundary for River Rch & Prof#=Elm Fork,ef5             , 1
Up Type= 0
Dn Type= 0
Boundary for River Rch & Prof#=Elm Fork,ef4             , 1
Up Type= 0
Dn Type= 0
Boundary for River Rch & Prof#=Elm Fork,ef3             , 1
Up Type= 0
Dn Type= 0
Boundary for River Rch & Prof#=Elm Fork,PGBT split west , 1
Up Type= 0
Dn Type= 0
Boundary for River Rch & Prof#=Elm Fork,PGBT split east , 1
Up Type= 0
Dn Type= 0
Boundary for River Rch & Prof#=Elm Fork,ef3 ds          , 1
Up Type= 0
Dn Type= 1
Dn Known WS=428.77
Boundary for River Rch & Prof#=Elm Fork L-Spill,efl             , 1
Up Type= 3
Up Slope=0.0022
Dn Type= 0
Boundary for River Rch & Prof#=Elm Fork Split2,efs2            , 1
Up Type= 0
Dn Type= 0
Boundary for River Rch & Prof#=Main Stem,ms              , 1
Up Type= 0
Dn Type= 1
Dn Known WS=399.43
Boundary for River Rch & Prof#=West Fork,wf              , 1
Up Type= 0
Dn Type= 0
DSS Import GetInterval= 0
DSS Import GetPeak= 0
DSS Import FillOption= 0

--- CDC_Consolidated_Model.f03 (steady flow) ---

Flow Title=Exist: 10%,4%,2%,1%,0.2%,1%+ AEP [WF/CF]
Program Version=6.60
BEGIN FILE DESCRIPTION:
Existing: 10%, 4%, 2%, 1%, 0.2%, 1%+ ACE (Annual Exceedance Probability) peak flows
END FILE DESCRIPTION:
Number of Profiles= 6
Profile Names=10% AEP,4% AEP,2% AEP,1% AEP,0.2% AEP,1%+ AEP
River Rch & RM=Clear Fork,cf              ,64970
    6000    6000    7500   13000   46000   20000
River Rch & RM=Clear Fork,cf              ,40758
 16888.2 24229.7 30150.4 36439.7 47829.2   51898
River Rch & RM=Clear Fork,cf              ,34851
 18073.6 25728.1 32607.5 39595.5 55422.5   56561
River Rch & RM=Clear Fork,cf              ,8301
 18177.2 25697.1 32098.5   38676 55341.6   53426
River Rch & RM=West Fork,wf4             ,306141
 14492.1 23277.1 28328.4 34713.6 53773.235312.54
River Rch & RM=West Fork,wf4             ,256421
 14485.7 23242.7 28296.8 34679.9 53705.8 46599.4
River Rch & RM=West Fork,wf3             ,253939
   24811 37079.1 47142.2 56387.5 93008.669998.16
River Rch & RM=West Fork,wf3             ,247864
 24765.9   36988 47019.8   56328 93033.778339.77
River Rch & RM=West Fork,wf3             ,241937
 26078.6   38380 48806.5 58454.1 97222.368799.78
River Rch & RM=West Fork,wf3             ,234374
 27459.5 39495.3 50128.1 58970.5 99303.779600.89
River Rch & RM=West Fork,wf3             ,221540
 37501.5 53043.7 65417.7 75911.2119507.2115555.9
River Rch & RM=West Fork,wf3             ,208050
 30114.7 45467.8 57609.2 68793.5110744.7103320.5
Boundary for River Rch & Prof#=Clear Fork,cf              , 1
Up Type= 0
Dn Type= 0
Boundary for River Rch & Prof#=Clear Fork,cf              , 2
Up Type= 0
Dn Type= 0
Boundary for River Rch & Prof#=Clear Fork,cf              , 3
Up Type= 0
Dn Type= 0
Boundary for River Rch & Prof#=Clear Fork,cf              , 4
Up Type= 0
Dn Type= 0
Boundary for River Rch & Prof#=Clear Fork,cf              , 5
Up Type= 0
Dn Type= 0
Boundary for River Rch & Prof#=Clear Fork,cf              , 6
Up Type= 0
Dn Type= 0
Boundary for River Rch & Prof#=West Fork,wf4             , 1
Up Type= 0
Dn Type= 0
Boundary for River Rch & Prof#=West Fork,wf4             , 2
Up Type= 0
Dn Type= 0
Boundary for River Rch & Prof#=West Fork,wf4             , 3
Up Type= 0
Dn Type= 0
Boundary for River Rch & Prof#=West Fork,wf4             , 4
Up Type= 0
Dn Type= 0
Boundary for River Rch & Prof#=West Fork,wf4             , 5
Up Type= 0
Dn Type= 0
Boundary for River Rch & Prof#=West Fork,wf4             , 6
Up Type= 0
Dn Type= 0
Boundary for River Rch & Prof#=West Fork,wf3             , 1
Up Type= 0
Dn Type= 1
Dn Known WS=506.23
Boundary for River Rch & Prof#=West Fork,wf3             , 2
Up Type= 0
Dn Type= 1
Dn Known WS=509.09
Boundary for River Rch & Prof#=West Fork,wf3             , 3
Up Type= 0
Dn Type= 1
Dn Known WS=510.88
Boundary for River Rch & Prof#=West Fork,wf3             , 4
Up Type= 0
Dn Type= 1
Dn Known WS=512.34
Boundary for River Rch & Prof#=West Fork,wf3             , 5
Up Type= 0
Dn Type= 1
Dn Known WS=516.61
Boundary for River Rch & Prof#=West Fork,wf3             , 6
Up Type= 0
Dn Type= 1
Dn Known WS=516.36
Set Internal Change=Clear Fork      ,cf              ,43004   , 6 , 3 ,611.2
Observed RC=Fort Worth Gage,West Fork       ,wf3             ,251524.5,0
Observed RC Desc=Data from USGS June 2007
Observed RC Data= 14
  519.54       0     520      24     521     923     522    2710     523    5550
     524    9310     525   13600     526   18400     527   23500     528   29100
     529   35200   529.1   35900   529.2   36500  529.24   36800
Observed RC Point Data= 0
Observed RC=Clear Fork Gage,Clear Fork      ,cf              ,12901.55,0
Observed RC Desc=Data from USGS June 2007
Observed RC Data= 24
  540.97       0     541     .06   541.5      23     542     207   542.5     767
     543    1350   543.5    2080     544    3030   544.5    4150     545    5430
   545.5    6850     546    8310   546.5    9800     547   11400   547.5   13000
     548   14700   548.5   16400     549   18200   549.5   20100   549.6   20500
   549.7   20900   549.8   21300   549.9   21700  549.91   21700
Observed RC Point Data= 0
DSS Import GetInterval= 0
DSS Import GetPeak= 0
DSS Import FillOption= 0

--- CDC_Consolidated_Model.f04 (steady flow) ---

Flow Title=Exist: FEMA Floodway 1% AEP [WF/EF/TRMS]
Program Version=6.60
BEGIN FILE DESCRIPTION:
Existing: 1% ACE (Annual Exceedance Probability) peak flows
END FILE DESCRIPTION:
Number of Profiles= 2
Profile Names=1% AEP,1% AEP FW
River Rch & RM=Elm Fork,ef6             ,153340
    7000    7000
River Rch & RM=Elm Fork,ef5             ,147501
   21000   21000
River Rch & RM=Elm Fork,ef4             ,138526
    7000    7000
River Rch & RM=Elm Fork,ef3             ,125671
   21000   21000
River Rch & RM=Elm Fork,ef3             ,118745
   21000   21000
River Rch & RM=Elm Fork,ef3             ,112469
   21000   21000
River Rch & RM=Elm Fork,ef3             ,107977
   44597   44597
River Rch & RM=Elm Fork,ef3             ,102709
   43553   43553
River Rch & RM=Elm Fork,ef3             ,93155
   41276   41276
River Rch & RM=Elm Fork,ef3             ,80596
   43419   43419
River Rch & RM=Elm Fork,ef3             ,64635
   42825   42825
River Rch & RM=Elm Fork,ef3             ,53311
   42825   42825
River Rch & RM=Elm Fork,ef2             ,48931
   32000   32000
River Rch & RM=Elm Fork,ef1             ,31628
   42825   42825
River Rch & RM=Elm Fork,ef1             ,30779
   41462   41462
River Rch & RM=Elm Fork,ef1             ,24559
   41153   41153
River Rch & RM=Elm Fork,ef1             ,17640
   41366   41366
River Rch & RM=Elm Fork L-Spill,efl             ,15577
   21000   21000
River Rch & RM=Elm Fork Split1,efs1            ,9111
10824.8510824.85
River Rch & RM=Elm Fork Split2,efs2            ,133117
   14000   14000
River Rch & RM=Main Stem,ms              ,148139
  118755  118755
River Rch & RM=Main Stem,ms              ,110079
  113234  113234
River Rch & RM=Main Stem,ms              ,82348
  118845  118845
River Rch & RM=Main Stem,ms              ,76808
  117706  117706
River Rch & RM=Main Stem,ms              ,53576
  117706  117706
River Rch & RM=Main Stem,ms              ,51043
  117706  117706
River Rch & RM=West Fork,wf3             ,206158
   68794   68794
River Rch & RM=West Fork,wf3             ,184441
   86097   86097
River Rch & RM=West Fork,wf3             ,162387
   82295   82295
River Rch & RM=West Fork,wf3             ,140843
   97693   97693
River Rch & RM=West Fork,wf3             ,133374
   95167   95167
River Rch & RM=West Fork,wf3             ,123707
   96559   96559
River Rch & RM=West Fork,wf3             ,116017
   95854   95854
River Rch & RM=West Fork,wf3f            ,112687
   47926   47926
River Rch & RM=West Fork,wf3e            ,111697
   47928   47928
River Rch & RM=West Fork,wf3d            ,107732
   95854   95854
River Rch & RM=West Fork,wf3d            ,96217
   93111   93111
River Rch & RM=West Fork,wf3b            ,84526
   49000   49000
River Rch & RM=West Fork,wf3c            ,80116
   44111   44111
River Rch & RM=West Fork,wf3a            ,74827
   93111   93111
River Rch & RM=West Fork,wf2             ,53716
   86111   86111
River Rch & RM=West Fork,wf2             ,35195
   84997   84997
River Rch & RM=West Fork,wf1             ,34256
   91997   91997
River Rch & RM=West Fork,wf1             ,24876
   95062   95062
River Rch & RM=West Fork,wf1             ,11909
   94443   94443
River Rch & RM=West Fork,wf1             ,1494
   93993   93993
River Rch & RM=West Fork Split,wfs             ,56034
    7000    7000
Boundary for River Rch & Prof#=Elm Fork,ef6             , 1
Up Type= 3
Up Slope=0.001
Dn Type= 0
Boundary for River Rch & Prof#=Elm Fork,ef6             , 2
Up Type= 3
Up Slope=0.001
Dn Type= 0
Boundary for River Rch & Prof#=Elm Fork,ef5             , 1
Up Type= 0
Dn Type= 0
Boundary for River Rch & Prof#=Elm Fork,ef5             , 2
Up Type= 0
Dn Type= 0
Boundary for River Rch & Prof#=Elm Fork,ef4             , 1
Up Type= 0
Dn Type= 0
Boundary for River Rch & Prof#=Elm Fork,ef4             , 2
Up Type= 0
Dn Type= 0
Boundary for River Rch & Prof#=Elm Fork,ef3             , 1
Up Type= 0
Dn Type= 0
Boundary for River Rch & Prof#=Elm Fork,ef3             , 2
Up Type= 0
Dn Type= 0
Boundary for River Rch & Prof#=Elm Fork,ef2             , 1
Up Type= 0
Dn Type= 0
Boundary for River Rch & Prof#=Elm Fork,ef2             , 2
Up Type= 0
Dn Type= 0
Boundary for River Rch & Prof#=Elm Fork,ef1             , 1
Up Type= 0
Dn Type= 0
Boundary for River Rch & Prof#=Elm Fork,ef1             , 2
Up Type= 0
Dn Type= 0
Boundary for River Rch & Prof#=Elm Fork L-Spill,efl             , 1
Up Type= 3
Up Slope=0.0022
Dn Type= 0
Boundary for River Rch & Prof#=Elm Fork L-Spill,efl             , 2
Up Type= 3
Up Slope=0.0022
Dn Type= 0
Boundary for River Rch & Prof#=Elm Fork Split1,efs1            , 1
Up Type= 0
Dn Type= 0
Boundary for River Rch & Prof#=Elm Fork Split1,efs1            , 2
Up Type= 0
Dn Type= 0
Boundary for River Rch & Prof#=Elm Fork Split2,efs2            , 1
Up Type= 0
Dn Type= 0
Boundary for River Rch & Prof#=Elm Fork Split2,efs2            , 2
Up Type= 0
Dn Type= 0
Boundary for River Rch & Prof#=Main Stem,ms              , 1
Up Type= 0
Dn Type= 1
Dn Known WS=394.69
Boundary for River Rch & Prof#=Main Stem,ms              , 2
Up Type= 0
Dn Type= 1
Dn Known WS=394.69
Boundary for River Rch & Prof#=West Fork,wf3             , 1
Up Type= 0
Dn Type= 0
Boundary for River Rch & Prof#=West Fork,wf3             , 2
Up Type= 0
Dn Type= 0
Boundary for River Rch & Prof#=West Fork,wf3f            , 1
Up Type= 0
Dn Type= 0
Boundary for River Rch & Prof#=West Fork,wf3f            , 2
Up Type= 0
Dn Type= 0
Boundary for River Rch & Prof#=West Fork,wf3e            , 1
Up Type= 0
Dn Type= 0
Boundary for River Rch & Prof#=West Fork,wf3e            , 2
Up Type= 0
Dn Type= 0
Boundary for River Rch & Prof#=West Fork,wf3d            , 1
Up Type= 0
Dn Type= 0
Boundary for River Rch & Prof#=West Fork,wf3d            , 2
Up Type= 0
Dn Type= 0
Boundary for River Rch & Prof#=West Fork,wf3b            , 1
Up Type= 0
Dn Type= 0
Boundary for River Rch & Prof#=West Fork,wf3b            , 2
Up Type= 0
Dn Type= 0
Boundary for River Rch & Prof#=West Fork,wf3c            , 1
Up Type= 0
Dn Type= 0
Boundary for River Rch & Prof#=West Fork,wf3c            , 2
Up Type= 0
Dn Type= 0
Boundary for River Rch & Prof#=West Fork,wf3a            , 1
Up Type= 0
Dn Type= 0
Boundary for River Rch & Prof#=West Fork,wf3a            , 2
Up Type= 0
Dn Type= 0
Boundary for River Rch & Prof#=West Fork,wf2             , 1
Up Type= 0
Dn Type= 0
Boundary for River Rch & Prof#=West Fork,wf2             , 2
Up Type= 0
Dn Type= 0
Boundary for River Rch & Prof#=West Fork,wf1             , 1
Up Type= 0
Dn Type= 0
Boundary for River Rch & Prof#=West Fork,wf1             , 2
Up Type= 0
Dn Type= 0
Boundary for River Rch & Prof#=West Fork Split,wfs             , 1
Up Type= 0
Dn Type= 0
Boundary for River Rch & Prof#=West Fork Split,wfs             , 2
Up Type= 0
Dn Type= 0
DSS Import GetInterval= 0
DSS Import GetPeak= 0
DSS Import FillOption= 0

--- CDC_Consolidated_Model.f05 (steady flow) ---

Flow Title=Exist: FEMA Floodway 1% AEP [WF/CF]
Program Version=6.60
BEGIN FILE DESCRIPTION:
Existing: 1% ACE (Annual Exceedance Probability) peak flows
END FILE DESCRIPTION:
Number of Profiles= 2
Profile Names=1% AEP,1% AEP FW
River Rch & RM=Clear Fork,cf              ,64970
   13000   13000
River Rch & RM=Clear Fork,cf              ,40758
 36439.7 36439.7
River Rch & RM=Clear Fork,cf              ,34851
 39595.5 39595.5
River Rch & RM=Clear Fork,cf              ,8301
   38676   38676
River Rch & RM=West Fork,wf4             ,306141
 34713.6 34713.6
River Rch & RM=West Fork,wf4             ,256421
 34679.9 34679.9
River Rch & RM=West Fork,wf3             ,253939
 56387.5 56387.5
River Rch & RM=West Fork,wf3             ,247864
   56328   56328
River Rch & RM=West Fork,wf3             ,241937
 58454.1 58454.1
River Rch & RM=West Fork,wf3             ,234374
 58970.5 58970.5
River Rch & RM=West Fork,wf3             ,221540
 75911.2 75911.2
River Rch & RM=West Fork,wf3             ,208050
 68793.5 68793.5
Boundary for River Rch & Prof#=Clear Fork,cf              , 1
Up Type= 0
Dn Type= 0
Boundary for River Rch & Prof#=Clear Fork,cf              , 2
Up Type= 0
Dn Type= 0
Boundary for River Rch & Prof#=West Fork,wf4             , 1
Up Type= 0
Dn Type= 0
Boundary for River Rch & Prof#=West Fork,wf4             , 2
Up Type= 0
Dn Type= 0
Boundary for River Rch & Prof#=West Fork,wf3             , 1
Up Type= 0
Dn Type= 1
Dn Known WS=512.34
Boundary for River Rch & Prof#=West Fork,wf3             , 2
Up Type= 0
Dn Type= 1
Dn Known WS=513.13
DSS Import GetInterval= 0
DSS Import GetPeak= 0
DSS Import FillOption= 0

--- CDC_Consolidated_Model.f06 (steady flow) ---

Flow Title=Exist: 1%+ AEP [WF/EF/TRMS]
Program Version=6.60
BEGIN FILE DESCRIPTION:
Existing: 1%+ ACE (Annual Exceedance Probability) peak flows
END FILE DESCRIPTION:
Number of Profiles= 1
Profile Names=1%+ AEP
River Rch & RM=Elm Fork,ef3             ,107977
   59842
River Rch & RM=Elm Fork,ef3             ,102709
   59842
River Rch & RM=Elm Fork,PGBT split west ,97191
   55000
River Rch & RM=Elm Fork,PGBT split east ,98000
    4842
River Rch & RM=Elm Fork,ef3 ds          ,87661
   59842
River Rch & RM=Elm Fork,ef3 ds          ,87553
   55341
River Rch & RM=Elm Fork,ef3 ds          ,80596
   59203
River Rch & RM=Elm Fork,ef3 ds          ,72731
   59203
River Rch & RM=Elm Fork,ef3 ds          ,53311
   59386
River Rch & RM=Elm Fork,ef3 ds          ,48931
   59386
River Rch & RM=Elm Fork,ef3 ds          ,31628
   56981
River Rch & RM=Elm Fork,ef3 ds          ,23599
   56321
River Rch & RM=Elm Fork,ef3 ds          ,18646
   56321
River Rch & RM=Main Stem,ms              ,148139
  173645
River Rch & RM=Main Stem,ms              ,110079
  164987
River Rch & RM=Main Stem,ms              ,82348
  167701
River Rch & RM=Main Stem,ms              ,76808
  167820
River Rch & RM=Main Stem,ms              ,53576
  167820
River Rch & RM=Main Stem,ms              ,51043
  167820
River Rch & RM=West Fork,wf              ,206158
  103321
River Rch & RM=West Fork,wf              ,184441
  145036
River Rch & RM=West Fork,wf              ,162387
  133941
River Rch & RM=West Fork,wf              ,140843
  156537
River Rch & RM=West Fork,wf              ,133374
  146694
River Rch & RM=West Fork,wf              ,123707
  149572
River Rch & RM=West Fork,wf              ,116017
  143489
River Rch & RM=West Fork,wf              ,107732
  143489
River Rch & RM=West Fork,wf              ,96217
  139766
River Rch & RM=West Fork,wf              ,74827
  139766
River Rch & RM=West Fork,wf              ,53716
  109000
River Rch & RM=West Fork,wf              ,35195
  135394
River Rch & RM=West Fork,wf              ,34256
  135394
River Rch & RM=West Fork,wf              ,24876
  156216
River Rch & RM=West Fork,wf              ,11909
  112739
River Rch & RM=West Fork,wf              ,1494
  138320
Boundary for River Rch & Prof#=Elm Fork,ef3             , 1
Up Type= 0
Dn Type= 0
Boundary for River Rch & Prof#=Elm Fork,PGBT split west , 1
Up Type= 0
Dn Type= 0
Boundary for River Rch & Prof#=Elm Fork,PGBT split east , 1
Up Type= 0
Dn Type= 0
Boundary for River Rch & Prof#=Elm Fork,ef3 ds          , 1
Up Type= 0
Dn Type= 1
Dn Known WS=428.77
Boundary for River Rch & Prof#=Main Stem,ms              , 1
Up Type= 0
Dn Type= 1
Dn Known WS=398.17
Boundary for River Rch & Prof#=West Fork,wf              , 1
Up Type= 0
Dn Type= 0
DSS Import GetInterval= 0
DSS Import GetPeak= 0
DSS Import FillOption= 0

--- CDC_Consolidated_Model.f12 (steady flow) ---

Flow Title=CDC: 50% to 1% AEP [WF/EF/TRMS]
Program Version=5.07
BEGIN FILE DESCRIPTION:
CDC: 50%, 20%, 10%, 4%, 2%, 1% ACE (Annual Exceedance Probability) peak flows
END FILE DESCRIPTION:
Number of Profiles= 6
Profile Names=50% AEP,20% AEP,10% AEP,4% AEP,2% AEP,1% AEP
River Rch & RM=Elm Fork,ef6             ,153328
    1800    2400    2700    3200    3700       1
River Rch & RM=Elm Fork,ef6             ,153092
    3200    4400    5400    6600    7700       1
River Rch & RM=Elm Fork,ef6             ,150592
    1600    2000    2300    2700    3100       1
River Rch & RM=Elm Fork,ef5             ,147489
    4900    6500    7600    9200   10500   21000
River Rch & RM=Elm Fork,ef5             ,144474
    2600    3300    3800    4500   10200   21000
River Rch & RM=Elm Fork,ef5             ,142900
    4200    5300    6100    7300   10200   21000
River Rch & RM=Elm Fork,ef4             ,139890
    3850    4840    5590    6750    9670   20330
River Rch & RM=Elm Fork,ef4             ,138514
    2400    2900    3000    3200    4000    7100
River Rch & RM=Elm Fork,ef3             ,125658
    4200    5300    6100    7300   10200   21000
River Rch & RM=Elm Fork,ef3             ,124975
    2800    4100    4800    5800   10200   21000
River Rch & RM=Elm Fork,ef3             ,118732
    6300    8100    9500   11500   14000   21000
River Rch & RM=Elm Fork,ef3             ,112732
    5900    7900    8900   11500   13500   21000
River Rch & RM=Elm Fork,ef3             ,110572
   10500   14500   17000   21500   26000   30500
River Rch & RM=Elm Fork,ef3             ,102686
   14500   23500   29000   35500   42000   49500
River Rch & RM=Elm Fork,ef3             ,93940
   13500   21000   26000   33000   40000   48000
River Rch & RM=Elm Fork,ef3             ,83530
   13000   20000   25000   31500   37500   45500
River Rch & RM=Elm Fork,ef3             ,80579
   13500   21000   26000   33000   38500   47000
River Rch & RM=Elm Fork,ef3             ,72713
   13500   20500   26500   33000   39000   47500
River Rch & RM=Elm Fork,ef3             ,71682
   13000   20500   26500   33000   38500   47000
River Rch & RM=Elm Fork,ef3             ,69701
   12500   20500   26500   33500   39000   47500
River Rch & RM=Elm Fork,ef3             ,67364
   12500   20500   26500   33500   39000   47500
River Rch & RM=Elm Fork,ef3             ,60810
   12500   20500   26500   33500   39500   48000
River Rch & RM=Elm Fork,ef3             ,57195
   12000   19500   25500   33000   39000   47000
River Rch & RM=Elm Fork,ef3             ,53292
   15500   20000   26500   34000   40000   48000
River Rch & RM=Elm Fork,ef2             ,48911
   14700   18700   24400   30500   34200   38200
River Rch & RM=Elm Fork,ef1             ,31605
   15500   20000   26500   34000   40000   48000
River Rch & RM=Elm Fork,ef1             ,30755
   11500   18500   24000   31000   37500   45000
River Rch & RM=Elm Fork,ef1             ,23574
   11500   18000   24000   31000   38000   45000
River Rch & RM=Elm Fork,ef1             ,21333
   11500   18000   23500   30500   37500   44500
River Rch & RM=Elm Fork,ef1             ,18621
   11500   18000   23500   31000   38000   45500
River Rch & RM=Elm Fork,ef1             ,12658
   11500   18000   23000   29500   37500   44500
River Rch & RM=Elm Fork L-Spill,efl2            ,20757
    2500    3400    4000    4800   10500   21000
River Rch & RM=Elm Fork L-Spill,efl1            ,1396
    1800    2650    3200    3800    6400    6800
River Rch & RM=Elm Fork Split1,efs1            ,9111
     800    1300    2100    3500    5800    9800
River Rch & RM=Elm Fork Split2,efs2            ,139902
       1       1       1       1       1    1320
River Rch & RM=Elm Fork Split2,efs2            ,132950
    1800    2400    3100    4100    6200   13900
River Rch & RM=L-Overflow,efs3            ,6082
       1       1       1     125    2200   10100
River Rch & RM=Main Stem,ms              ,148136
   24000   39500   55000   87000  110000  129000
River Rch & RM=Main Stem,ms              ,138046
   23500   38500   54000   86000  109000  129000
River Rch & RM=Main Stem,ms              ,91392
   23500   38500   54000   86000  109000  129000
River Rch & RM=Main Stem,ms              ,82361
   20000   33500   50500   79500  102000  124000
River Rch & RM=Main Stem,ms              ,77843
   24500   40000   54000   83500  107000  130000
River Rch & RM=Main Stem,ms              ,68027
   24500   40000   54000   83000  107000  130000
River Rch & RM=Main Stem,ms              ,51060
   23500   39000   53000   82000  105000  129000
River Rch & RM=West Fork,wf3             ,206218
   16500   28500   39500   55000   67000   78000
River Rch & RM=West Fork,wf3             ,184495
   18000   32500   47500   66500   79000   91500
River Rch & RM=West Fork,wf3             ,162435
   16500   30000   43500   62500   75500   89000
River Rch & RM=West Fork,wf3             ,140885
   20500   35500   50000   72500   89500  110000
River Rch & RM=West Fork,wf3             ,133413
   19500   34000   48000   70000   87000  108000
River Rch & RM=West Fork,wf3             ,123744
   19500   34000   48500   71000   88000  109000
River Rch & RM=West Fork,wf3             ,116053
   19000   33000   47500   70000   87500  108000
River Rch & RM=West Fork,wf3f            ,111680
       1    3600   13000   30000   43500   64500
River Rch & RM=West Fork,wf3e            ,111679
   18999   29400   34500   40000   44000   43500
River Rch & RM=West Fork,wf3d            ,107775
   19000   33000   47500   70000   87500  108000
River Rch & RM=West Fork,wf3d            ,96240
   18500   32000   46500   68500   85500  107000
River Rch & RM=West Fork,wf3b            ,84548
   13700   19000   25000   35500   43500   55500
River Rch & RM=West Fork,wf3c            ,84549
    4800   13000   21500   33000   42000   51500
River Rch & RM=West Fork,wf3a            ,74891
   18500   32000   46500   68500   85500  107000
River Rch & RM=West Fork,wf3a            ,70006
   18000   30500   45500   67500   84500  109000
River Rch & RM=West Fork,wf2             ,53730
   17500   30000   48000   69500   82100   91500
River Rch & RM=West Fork,wf1             ,34268
   17500   30000   48000   72500   90000  106000
River Rch & RM=West Fork,wf1             ,18823
   17500   28000   43500   67500   85500  103000
River Rch & RM=West Fork,wf1             ,11911
   17500   28000   44000   68500   86500  104000
River Rch & RM=West Fork,wf1             ,8149
   17000   28000   43000   67500   85500  103000
River Rch & RM=West Fork Split,wfs             ,56004
       1       1       1    3000    7900   14500
Boundary for River Rch & Prof#=Elm Fork,ef6             , 1
Up Type= 3
Up Slope=0.001
Dn Type= 0
Boundary for River Rch & Prof#=Elm Fork,ef6             , 2
Up Type= 3
Up Slope=0.001
Dn Type= 0
Boundary for River Rch & Prof#=Elm Fork,ef6             , 3
Up Type= 3
Up Slope=0.001
Dn Type= 0
Boundary for River Rch & Prof#=Elm Fork,ef6             , 4
Up Type= 3
Up Slope=0.001
Dn Type= 0
Boundary for River Rch & Prof#=Elm Fork,ef6             , 5
Up Type= 3
Up Slope=0.001
Dn Type= 0
Boundary for River Rch & Prof#=Elm Fork,ef6             , 6
Up Type= 3
Up Slope=0.001
Dn Type= 0
Boundary for River Rch & Prof#=Elm Fork,ef5             , 1
Up Type= 0
Dn Type= 0
Boundary for River Rch & Prof#=Elm Fork,ef5             , 2
Up Type= 0
Dn Type= 0
Boundary for River Rch & Prof#=Elm Fork,ef5             , 3
Up Type= 0
Dn Type= 0
Boundary for River Rch & Prof#=Elm Fork,ef5             , 4
Up Type= 0
Dn Type= 0
Boundary for River Rch & Prof#=Elm Fork,ef5             , 5
Up Type= 0
Dn Type= 0
Boundary for River Rch & Prof#=Elm Fork,ef5             , 6
Up Type= 0
Dn Type= 0
Boundary for River Rch & Prof#=Elm Fork,ef4             , 1
Up Type= 0
Dn Type= 0
Boundary for River Rch & Prof#=Elm Fork,ef4             , 2
Up Type= 0
Dn Type= 0
Boundary for River Rch & Prof#=Elm Fork,ef4             , 3
Up Type= 0
Dn Type= 0
Boundary for River Rch & Prof#=Elm Fork,ef4             , 4
Up Type= 0
Dn Type= 0
Boundary for River Rch & Prof#=Elm Fork,ef4             , 5
Up Type= 0
Dn Type= 0
Boundary for River Rch & Prof#=Elm Fork,ef4             , 6
Up Type= 0
Dn Type= 0
Boundary for River Rch & Prof#=Elm Fork,ef3             , 1
Up Type= 0
Dn Type= 0
Boundary for River Rch & Prof#=Elm Fork,ef3             , 2
Up Type= 0
Dn Type= 0
Boundary for River Rch & Prof#=Elm Fork,ef3             , 3
Up Type= 0
Dn Type= 0
Boundary for River Rch & Prof#=Elm Fork,ef3             , 4
Up Type= 0
Dn Type= 0
Boundary for River Rch & Prof#=Elm Fork,ef3             , 5
Up Type= 0
Dn Type= 0
Boundary for River Rch & Prof#=Elm Fork,ef3             , 6
Up Type= 0
Dn Type= 0
Boundary for River Rch & Prof#=Elm Fork,ef2             , 1
Up Type= 0
Dn Type= 0
Boundary for River Rch & Prof#=Elm Fork,ef2             , 2
Up Type= 0
Dn Type= 0
Boundary for River Rch & Prof#=Elm Fork,ef2             , 3
Up Type= 0
Dn Type= 0
Boundary for River Rch & Prof#=Elm Fork,ef2             , 4
Up Type= 0
Dn Type= 0
Boundary for River Rch & Prof#=Elm Fork,ef2             , 5
Up Type= 0
Dn Type= 0
Boundary for River Rch & Prof#=Elm Fork,ef2             , 6
Up Type= 0
Dn Type= 0
Boundary for River Rch & Prof#=Elm Fork,ef1             , 1
Up Type= 0
Dn Type= 0
Boundary for River Rch & Prof#=Elm Fork,ef1             , 2
Up Type= 0
Dn Type= 0
Boundary for River Rch & Prof#=Elm Fork,ef1             , 3
Up Type= 0
Dn Type= 0
Boundary for River Rch & Prof#=Elm Fork,ef1             , 4
Up Type= 0
Dn Type= 0
Boundary for River Rch & Prof#=Elm Fork,ef1             , 5
Up Type= 0
Dn Type= 0
Boundary for River Rch & Prof#=Elm Fork,ef1             , 6
Up Type= 0
Dn Type= 0
Boundary for River Rch & Prof#=Elm Fork L-Spill,efl2            , 1
Up Type= 0
Dn Type= 0
Boundary for River Rch & Prof#=Elm Fork L-Spill,efl2            , 2
Up Type= 0
Dn Type= 0
Boundary for River Rch & Prof#=Elm Fork L-Spill,efl2            , 3
Up Type= 0
Dn Type= 0
Boundary for River Rch & Prof#=Elm Fork L-Spill,efl2            , 4
Up Type= 0
Dn Type= 0
Boundary for River Rch & Prof#=Elm Fork L-Spill,efl2            , 5
Up Type= 0
Dn Type= 0
Boundary for River Rch & Prof#=Elm Fork L-Spill,efl2            , 6
Up Type= 0
Dn Type= 0
Boundary for River Rch & Prof#=Elm Fork L-Spill,efl1            , 1
Up Type= 0
Dn Type= 0
Boundary for River Rch & Prof#=Elm Fork L-Spill,efl1            , 2
Up Type= 0
Dn Type= 0
Boundary for River Rch & Prof#=Elm Fork L-Spill,efl1            , 3
Up Type= 0
Dn Type= 0
Boundary for River Rch & Prof#=Elm Fork L-Spill,efl1            , 4
Up Type= 0
Dn Type= 0
Boundary for River Rch & Prof#=Elm Fork L-Spill,efl1            , 5
Up Type= 0
Dn Type= 0
Boundary for River Rch & Prof#=Elm Fork L-Spill,efl1            , 6
Up Type= 0
Dn Type= 0
Boundary for River Rch & Prof#=Elm Fork Split1,efs1            , 1
Up Type= 0
Dn Type= 0
Boundary for River Rch & Prof#=Elm Fork Split1,efs1            , 2
Up Type= 0
Dn Type= 0
Boundary for River Rch & Prof#=Elm Fork Split1,efs1            , 3
Up Type= 0
Dn Type= 0
Boundary for River Rch & Prof#=Elm Fork Split1,efs1            , 4
Up Type= 0
Dn Type= 0
Boundary for River Rch & Prof#=Elm Fork Split1,efs1            , 5
Up Type= 0
Dn Type= 0
Boundary for River Rch & Prof#=Elm Fork Split1,efs1            , 6
Up Type= 0
Dn Type= 0
Boundary for River Rch & Prof#=Elm Fork Split2,efs2            , 1
Up Type= 0
Dn Type= 0
Boundary for River Rch & Prof#=Elm Fork Split2,efs2            , 2
Up Type= 0
Dn Type= 0
Boundary for River Rch & Prof#=Elm Fork Split2,efs2            , 3
Up Type= 0
Dn Type= 0
Boundary for River Rch & Prof#=Elm Fork Split2,efs2            , 4
Up Type= 0
Dn Type= 0
Boundary for River Rch & Prof#=Elm Fork Split2,efs2            , 5
Up Type= 0
Dn Type= 0
Boundary for River Rch & Prof#=Elm Fork Split2,efs2            , 6
Up Type= 0
Dn Type= 0
Boundary for River Rch & Prof#=L-Overflow,efs3            , 1
Up Type= 0
Dn Type= 0
Boundary for River Rch & Prof#=L-Overflow,efs3            , 2
Up Type= 0
Dn Type= 0
Boundary for River Rch & Prof#=L-Overflow,efs3            , 3
Up Type= 0
Dn Type= 0
Boundary for River Rch & Prof#=L-Overflow,efs3            , 4
Up Type= 0
Dn Type= 0
Boundary for River Rch & Prof#=L-Overflow,efs3            , 5
Up Type= 0
Dn Type= 0
Boundary for River Rch & Prof#=L-Overflow,efs3            , 6
Up Type= 0
Dn Type= 0
Boundary for River Rch & Prof#=Main Stem,ms              , 1
Up Type= 0
Dn Type= 1
Dn Known WS=378.4
Boundary for River Rch & Prof#=Main Stem,ms              , 2
Up Type= 0
Dn Type= 1
Dn Known WS=383.5
Boundary for River Rch & Prof#=Main Stem,ms              , 3
Up Type= 0
Dn Type= 1
Dn Known WS=386.58
Boundary for River Rch & Prof#=Main Stem,ms              , 4
Up Type= 0
Dn Type= 1
Dn Known WS=390.97
Boundary for River Rch & Prof#=Main Stem,ms              , 5
Up Type= 0
Dn Type= 1
Dn Known WS=393.46
Boundary for River Rch & Prof#=Main Stem,ms              , 6
Up Type= 0
Dn Type= 1
Dn Known WS=395.53
Boundary for River Rch & Prof#=West Fork,wf3             , 1
Up Type= 0
Dn Type= 0
Boundary for River Rch & Prof#=West Fork,wf3             , 2
Up Type= 0
Dn Type= 0
Boundary for River Rch & Prof#=West Fork,wf3             , 3
Up Type= 0
Dn Type= 0
Boundary for River Rch & Prof#=West Fork,wf3             , 4
Up Type= 0
Dn Type= 0
Boundary for River Rch & Prof#=West Fork,wf3             , 5
Up Type= 0
Dn Type= 0
Boundary for River Rch & Prof#=West Fork,wf3             , 6
Up Type= 0
Dn Type= 0
Boundary for River Rch & Prof#=West Fork,wf3f            , 1
Up Type= 0
Dn Type= 0
Boundary for River Rch & Prof#=West Fork,wf3f            , 2
Up Type= 0
Dn Type= 0
Boundary for River Rch & Prof#=West Fork,wf3f            , 3
Up Type= 0
Dn Type= 0
Boundary for River Rch & Prof#=West Fork,wf3f            , 4
Up Type= 0
Dn Type= 0
Boundary for River Rch & Prof#=West Fork,wf3f            , 5
Up Type= 0
Dn Type= 0
Boundary for River Rch & Prof#=West Fork,wf3f            , 6
Up Type= 0
Dn Type= 0
Boundary for River Rch & Prof#=West Fork,wf3e            , 1
Up Type= 0
Dn Type= 0
Boundary for River Rch & Prof#=West Fork,wf3e            , 2
Up Type= 0
Dn Type= 0
Boundary for River Rch & Prof#=West Fork,wf3e            , 3
Up Type= 0
Dn Type= 0
Boundary for River Rch & Prof#=West Fork,wf3e            , 4
Up Type= 0
Dn Type= 0
Boundary for River Rch & Prof#=West Fork,wf3e            , 5
Up Type= 0
Dn Type= 0
Boundary for River Rch & Prof#=West Fork,wf3e            , 6
Up Type= 0
Dn Type= 0
Boundary for River Rch & Prof#=West Fork,wf3d            , 1
Up Type= 0
Dn Type= 0
Boundary for River Rch & Prof#=West Fork,wf3d            , 2
Up Type= 0
Dn Type= 0
Boundary for River Rch & Prof#=West Fork,wf3d            , 3
Up Type= 0
Dn Type= 0
Boundary for River Rch & Prof#=West Fork,wf3d            , 4
Up Type= 0
Dn Type= 0
Boundary for River Rch & Prof#=West Fork,wf3d            , 5
Up Type= 0
Dn Type= 0
Boundary for River Rch & Prof#=West Fork,wf3d            , 6
Up Type= 0
Dn Type= 0
Boundary for River Rch & Prof#=West Fork,wf3b            , 1
Up Type= 0
Dn Type= 0
Boundary for River Rch & Prof#=West Fork,wf3b            , 2
Up Type= 0
Dn Type= 0
Boundary for River Rch & Prof#=West Fork,wf3b            , 3
Up Type= 0
Dn Type= 0
Boundary for River Rch & Prof#=West Fork,wf3b            , 4
Up Type= 0
Dn Type= 0
Boundary for River Rch & Prof#=West Fork,wf3b            , 5
Up Type= 0
Dn Type= 0
Boundary for River Rch & Prof#=West Fork,wf3b            , 6
Up Type= 0
Dn Type= 0
Boundary for River Rch & Prof#=West Fork,wf3c            , 1
Up Type= 0
Dn Type= 0
Boundary for River Rch & Prof#=West Fork,wf3c            , 2
Up Type= 0
Dn Type= 0
Boundary for River Rch & Prof#=West Fork,wf3c            , 3
Up Type= 0
Dn Type= 0
Boundary for River Rch & Prof#=West Fork,wf3c            , 4
Up Type= 0
Dn Type= 0
Boundary for River Rch & Prof#=West Fork,wf3c            , 5
Up Type= 0
Dn Type= 0
Boundary for River Rch & Prof#=West Fork,wf3c            , 6
Up Type= 0
Dn Type= 0
Boundary for River Rch & Prof#=West Fork,wf3a            , 1
Up Type= 0
Dn Type= 0
Boundary for River Rch & Prof#=West Fork,wf3a            , 2
Up Type= 0
Dn Type= 0
Boundary for River Rch & Prof#=West Fork,wf3a            , 3
Up Type= 0
Dn Type= 0
Boundary for River Rch & Prof#=West Fork,wf3a            , 4
Up Type= 0
Dn Type= 0
Boundary for River Rch & Prof#=West Fork,wf3a            , 5
Up Type= 0
Dn Type= 0
Boundary for River Rch & Prof#=West Fork,wf3a            , 6
Up Type= 0
Dn Type= 0
Boundary for River Rch & Prof#=West Fork,wf2             , 1
Up Type= 0
Dn Type= 0
Boundary for River Rch & Prof#=West Fork,wf2             , 2
Up Type= 0
Dn Type= 0
Boundary for River Rch & Prof#=West Fork,wf2             , 3
Up Type= 0
Dn Type= 0
Boundary for River Rch & Prof#=West Fork,wf2             , 4
Up Type= 0
Dn Type= 0
Boundary for River Rch & Prof#=West Fork,wf2             , 5
Up Type= 0
Dn Type= 0
Boundary for River Rch & Prof#=West Fork,wf2             , 6
Up Type= 0
Dn Type= 0
Boundary for River Rch & Prof#=West Fork,wf1             , 1
Up Type= 0
Dn Type= 0
Boundary for River Rch & Prof#=West Fork,wf1             , 2
Up Type= 0
Dn Type= 0
Boundary for River Rch & Prof#=West Fork,wf1             , 3
Up Type= 0
Dn Type= 0
Boundary for River Rch & Prof#=West Fork,wf1             , 4
Up Type= 0
Dn Type= 0
Boundary for River Rch & Prof#=West Fork,wf1             , 5
Up Type= 0
Dn Type= 0
Boundary for River Rch & Prof#=West Fork,wf1             , 6
Up Type= 0
Dn Type= 0
Boundary for River Rch & Prof#=West Fork Split,wfs             , 1
Up Type= 0
Dn Type= 0
Boundary for River Rch & Prof#=West Fork Split,wfs             , 2
Up Type= 0
Dn Type= 0
Boundary for River Rch & Prof#=West Fork Split,wfs             , 3
Up Type= 0
Dn Type= 0
Boundary for River Rch & Prof#=West Fork Split,wfs             , 4
Up Type= 0
Dn Type= 0
Boundary for River Rch & Prof#=West Fork Split,wfs             , 5
Up Type= 0
Dn Type= 0
Boundary for River Rch & Prof#=West Fork Split,wfs             , 6
Up Type= 0
Dn Type= 0
Set Internal Change=West Fork       ,wf2             ,41697   , 2 , 3 ,436.1
Set Internal Change=West Fork       ,wf2             ,37866   , 2 , 3 ,434.25
DSS Import GetInterval= 0
DSS Import GetPeak= 0
DSS Import FillOption= 0
