HEC-RAS study CDC_Consolidated_Model.prj: Upper Trinity CDC Consolidated Model

--- CDC_Consolidated_Model.g11 (geometry) --- (continued)

Type RM Length L Ch R = 3 ,39980   ,,,
BEGIN DESCRIPTION:
SH 183/Southwest Boulevard
Bridge data from 1975 survey.  Minimum low chord elev. 614.77.  Bridge width 85 feet.
Channel data from 1975 USACE field survey.
END DESCRIPTION:
Node Name=SH 183
Bridge Culvert--1,0,-1,-1, 0
Deck Dist Width WeirC Skew NumUp NumDn MinLoCord MaxHiCord MaxSubmerge Is_Ogee
7.5,85,2.6,0, 22, 22, , , 0.95, 0, 0,0,,
  1001.8 1098.75 1101.25    1106    1161  1163.5    1205    1223  1225.5  1285.5
    1288 1346.75 1349.25    1399  1401.5    1471  1473.5    1594  1596.5    1644
  1646.5  1693.4
  622.17   621.7  621.68  621.66  621.37  621.35  621.14  621.05  621.04  620.77
  620.76  620.48  620.46  620.22  620.21  619.83  619.82   619.2  619.19  618.62
  618.59     618
  618.37  617.96  617.95  617.93  617.64  617.63  617.42  617.33  617.31     617
  616.99  616.69  616.68  616.42  616.41  616.05  616.04  615.42   615.4  614.81
  614.77  614.35
  1001.8 1098.75 1101.25    1106    1161  1163.5    1205    1223  1225.5  1285.5
    1288 1346.75 1349.25    1399  1401.5    1471  1473.5    1594  1596.5    1644
  1646.5  1693.4
  622.17   621.7  621.68  621.66  621.37  621.35  621.14  621.05  621.04  620.77
  620.76  620.48  620.46  620.22  620.21  619.83  619.82   619.2  619.19  618.62
  618.59     618
  618.37  617.96  617.95  617.93  617.64  617.63  617.42  617.33  617.31     617
  616.99  616.69  616.68  616.42  616.41  616.05  616.04  615.42   615.4  614.81
  614.77  614.35
Pier Skew, UpSta & Num, DnSta & Num=  ,1100, 2 ,1100, 2 , 0 , 0 , 0 ,,
     2.5     2.5
     600     620
     2.5     2.5
     600     620
Pier Skew, UpSta & Num, DnSta & Num=  ,1162.25, 2 ,1162.25, 2 , 0 , 0 , 0 ,,
     2.5     2.5
     570     620
     2.5     2.5
     570     620
Pier Skew, UpSta & Num, DnSta & Num=  ,1224.25, 2 ,1224.25, 2 , 0 , 0 , 0 ,,
     2.5     2.5
     570     620
     2.5     2.5
     570     620
Pier Skew, UpSta & Num, DnSta & Num=  ,1286.75, 2 ,1286.75, 2 , 0 , 0 , 0 ,,
     2.5     2.5
     570     620
     2.5     2.5
     570     620
Pier Skew, UpSta & Num, DnSta & Num=  ,1348, 2 ,1348, 2 , 0 , 0 , 0 ,,
     2.5     2.5
     570     620
     2.5     2.5
     570     620
Pier Skew, UpSta & Num, DnSta & Num=  ,1400.25, 2 ,1400.25, 2 , 0 , 0 , 0 ,,
     2.5     2.5
     570     619
     2.5     2.5
     570     619
Pier Skew, UpSta & Num, DnSta & Num=  ,1472.25, 2 ,1472.25, 2 , 0 , 0 , 0 ,,
     2.5     2.5
     570     619
     2.5     2.5
     570     619
Pier Skew, UpSta & Num, DnSta & Num=  ,1645.25, 2 ,1645.25, 2 , 0 , 0 , 0 ,,
     2.5     2.5
     570     618
     2.5     2.5
     570     618
BR Coef=-1 , 0 , 0 ,1.05, 0 ,,,0.8,-1,0.5,1,
WSPro=,,,, 1 ,,,, 0 ,,,, 0 ,,,,-1 ,-1 ,-1 , 0 , 0 , 0 , 0 , 0
BC Design=,, 0 ,, 0 ,,,,,,
BC HTab HWMax=622.17
BC Use User HTab Curves=0
BC User HTab FreeFlow(D)= 0

Type RM Length L Ch R = 1 ,39929   ,95.9,96.3,99.7
BEGIN DESCRIPTION:
This cross section corresponds to cross section 39977 of the non-georeferenced CDC model which was the source of this model.
Duplication of following bridge cross-section without bridge piers.
Upstream end of Fort Worth Floodway.
Channel data from 1975 USACE field survey.
END DESCRIPTION:
XS GIS Cut Line= 2
2299248.380017766938253.76990765 2299703.3820877 6937732.9208633
#Sta/Elev= 30
  1001.8  622.17  1001.8   617.3    1037   600.9    1050   602.9    1058   601.9
    1072   601.9 1101.25   603.7    1106   603.5    1129   599.2    1157   597.4
    1175   590.6    1184   583.4    1191     580    1223     579    1232   583.4
    1240   584.1  1285.5   584.6    1303   584.6    1318   581.4    1337   580.4
    1396   580.7  1401.5   585.9    1458   588.5    1471   594.9  1473.5   597.8
    1480   602.2    1532   602.4    1644   600.5    1665   602.4  1693.4     618
#Mann= 3 ,0,0
  1001.8     .06       0    1157    .035       0    1480     .06       0
Bank Sta=1157,1480
XS Rating Curve= 0 ,0
Exp/Cntr=0.5,0.3

Type RM Length L Ch R = 1 ,39833   ,538.1,496.5,474.4
BEGIN DESCRIPTION:
This cross section corresponds to cross section 39879 of the non-georeferenced CDC model which was the source of this model.
Cross-section modified by USACE February 2007.  Effective  in LOB set at sta 2050, in ROB set at sta 2800.
99 feet downstream of S.H. 183 - Southwest Boulevard.
Channel data from 1975 USACE field survey.
END DESCRIPTION:
XS GIS Cut Line= 5
   2298618.45398   6939119.50899   2298788.15213   6938925.26889
   2299301.79513   6938337.33601   2299792.84107    6937775.2269
 2300025.2667818 6937509.5644535
#Sta/Elev= 30
    1000   618.6    1304   618.1    1319   619.5    1738     628    1875   622.9
    1901     623    1969   619.5    2038     615    2081   610.2    2157   605.3
    2180   604.7    2222   597.6    2283   595.3    2321     583 2343.81     582
 2370.81   578.8 2456.81   578.8 2482.81     582    2506   582.5    2519   585.6
    2585     588    2638   601.2    2700     601    2765   602.2    2786   603.8
    2791   602.3    2845   602.7    2904   603.6    3022   607.3    3138   608.2
#Mann= 3 ,0,0
    1000     .06       0    2157    .035       0    2786     .06       0
#XS Ineff= 4 ,-1
    1000    2050     610    2050    2157   605.3    2786    2800   603.8
    2800    3138     610
Permanent Ineff=
       F       F       F       F
Bank Sta=2157,2786
XS Rating Curve= 0 ,0
Exp/Cntr=0.3,0.1

Type RM Length L Ch R = 1 ,39337   ,320,280,247
BEGIN DESCRIPTION:
This cross section corresponds to cross section 39380 of the non-georeferenced CDC model which was the source of this model.
Cross-section modified by USACE February 2007.  Effective  in LOB set at sta 1580, in ROB set at sta 2450.  Old river channel in ROB.  Channel data from 1975 USACE field survey.
Note:  Channel dam indicated on 1991 topography has been removed by the TRWD after construction of the new downstream channel dam and during the completion of the original CDC Model.
END DESCRIPTION:
XS GIS Cut Line= 3
   2299575.70305   6939144.79109   2300039.24313   6938178.48396
    2300375.7546   6937120.47394
#Sta/Elev= 30
    1000     608    1167     607    1227   607.5    1363   605.6    1694   605.1
    1763   603.7    1773   603.4    1822   578.3    1849   578.6    1882   576.2
    1983   576.2    1994   577.7    2069   608.7    2097   609.2    2147   592.2
    2161   592.7    2180   588.6    2187   588.2    2224   592.6    2319   608.5
    2386   609.3    2415   608.5    2447   601.9    2537   603.6    2669   601.7
    2802     604    2902   603.8    2994   605.2    3079   603.6    3182   604.7
#Mann= 3 ,0,0
    1000     .06       0    1763    .035       0    2069     .06       0
#XS Ineff= 2 , 0
            1580     610    2450             610
Permanent Ineff=
       F       F
#Block Obstruct= 1 ,-1
    2097    2319   608.5
Bank Sta=1763,2069
XS Rating Curve= 0 ,0
Exp/Cntr=0.3,0.1

Type RM Length L Ch R = 1 ,39057   ,58,58,58
XS GIS Cut Line= 4
  2299479.566364 6940803.2307766 2300183.0383354 6938775.8264183
      2300405.25      6937290.92       2300429.4     6937142.698
#Sta/Elev= 30
  1009.4     622  1041.3     610    1091     610  1134.8     608  1243.6     604
  1340.3     602  2140.2     602  2345.8     604  2400.2     604  2661.8     602
  2823.7     602  2971.9     604  3478.3     602  3545.3     580  3562.8     578
  3572.1     576    3593   574.4    3643   574.4  3688.7     578  3698.8     580
  3705.5     582  3759.8     602  3960.1     602  4008.4     582  4068.4     582
  4114.7     598  4125.3     602    4407     602    4650     604    4807     604
#Mann= 3 ,0,0
  1009.4     .06       0  3478.3    .035       0  3759.8     .06       0
#XS Ineff= 5 ,-1
  1009.4    2150     602    2150    3300     610    3300  3478.3     602
  3759.8    4260     602    4260    4807     610
Permanent Ineff=
       F       F       F       F       F
#Block Obstruct= 1 ,-1
 3960.12  4125.3     602
Bank Sta=3478.3,3759.8
XS Rating Curve= 0 ,0
Exp/Cntr=0.3,0.1

Type RM Length L Ch R = 5 ,39006   ,,,
BEGIN DESCRIPTION:
Cityview Dam
Data from plans.  Crest elevation 585.4, width 12 feet.
END DESCRIPTION:
Node Name=Cityview Dam
IW Pilot Flow=0
#Inline Weir SE= 2
    3000   585.4    4000   585.4
IW Dist,WD,Coef,Skew,MaxSub,Min_El,Is_Ogee,SpillHt,DesHd
33,12,3,0,0.95,, 0 ,,,2,2,
Inline Weir Flap Gates= 0
IW Outlet Rating Curve= 0 ,False,,

Type RM Length L Ch R = 1 ,38999   ,17.7,16.8,16.3
BEGIN DESCRIPTION:
This cross section corresponds to cross section 39055 of the non-georeferenced CDC model which was the source of this model.
One-foot downstream of Cityview Dam.
Cross-section modified by USACE February 2007.
Ineffective flow in LOB due to group of structures, effective flow in ROB set at sta 4260.
Old river channel in ROB.
Channel data from 1975 USACE field survey.
END DESCRIPTION:
XS GIS Cut Line= 4
2299524.272482346940850.03415726   2300240.39496   6938786.17107
   2300421.66396   6937574.60689      2300474.54      6937190.25
#Sta/Elev= 30
  1009.4     622  1041.3     610    1091     610  1243.6     604  1340.3     602
  2140.2     602  2345.8     604  2661.8     602  2823.7     602  2971.9     604
  3478.3     602    3527     586  3533.1   585.4  3539.2     582  3545.3     580
  3572.1     576    3593   574.4    3643   574.4  3688.7     578  3705.5     582
  3711.2   585.4  3716.8     586  3759.8     602  3960.1     602  4008.4     582
  4068.4     582  4125.3     602    4407     602    4650     604    4807     604
#Mann= 3 ,0,0
  1009.4     .06       0  3478.3    .035       0  3759.8     .06       0
#XS Ineff= 5 ,-1
  1009.4    2150     602    2150    3300     610    3300  3478.3     602
  3759.8    4260     602    4260    4807     610
Permanent Ineff=
       F       F       F       F       F
#Block Obstruct= 1 ,-1
 3960.12  4125.3     602
Bank Sta=3478.3,3759.8
XS Rating Curve= 0 ,0
Exp/Cntr=0.3,0.1

Type RM Length L Ch R = 1 ,38982   ,285.9,287.5,291
BEGIN DESCRIPTION:
This cross section corresponds to cross section 39023 of the non-georeferenced CDC model which was the source of this model.
Cross-section modified by USACE February 2007.
39 feet downstream of Cityview Dam.  Ineffective flow in LOB due to group of structures, effective flow in ROB set at sta 4260.
Old river channel in ROB.
Channel data from 1975 USACE field survey.
END DESCRIPTION:
XS GIS Cut Line= 4
2299530.905865176940852.77955862      2299570.13      6940774.24
 2300259.3457513 6938788.5749798      2300487.99      6937196.98
#Sta/Elev= 30
  1009.4     622  1041.3     610    1091     610  1134.8     608  1243.6     604
  1340.3     602  2140.2     602  2345.8     604  2400.2     604  2661.8     602
  2823.7     602  2971.9     604  3478.3     602  3545.3     580  3562.8     578
  3572.1     576    3593   574.4    3643   574.4  3688.7     578  3698.8     580
  3705.5     582  3759.8     602  3960.1     602  4008.4     582  4068.4     582
  4114.7     598  4125.3     602    4407     602    4650     604    4807     604
#Mann= 3 ,0,0
  1009.4     .06       0  3478.3    .035       0  3759.8     .06       0
#XS Ineff= 5 ,-1
  1009.4    2150     602    2150    3300     610    3300  3478.3     602
  3759.8    4260     602    4260    4807     610
Permanent Ineff=
       F       F       F       F       F
#Block Obstruct= 1 ,-1
 3960.12  4125.3     602
Bank Sta=3478.3,3759.8
XS Rating Curve= 0 ,0
Exp/Cntr=0.3,0.1

Type RM Length L Ch R = 1 ,38695   ,574.5,636,683.1
BEGIN DESCRIPTION:
This cross section corresponds to cross section 38738 of the non-georeferenced CDC model which was the source of this model.
Cross-section modified by USACE February 2007.
Ineffective flow in LOB due to group of structures, effective flow in ROB set at sta 4290.
Old river channel in ROB.
Channel data from 1975 USACE field survey.
END DESCRIPTION:
XS GIS Cut Line= 3
   2299505.98206   6940902.74689   2300516.75005   6938938.63894
   2300862.11911   6936859.02007
#Sta/Elev= 30
    1000   623.5    1040   609.6    1078   611.3    1412   600.7    2223     601
    2240   604.6    2554   599.4    2605   602.1    2738   599.9    2859   603.5
    2951   601.3    3123   603.5    3583   600.6 3673.51   574.4 3726.51   574.4
    3792     579    3864     600    4099   601.3    4155   581.2    4207   581.2
    4251   599.8    4398   600.9    4473   597.8    4524   601.9    4592   601.8
    4626   598.4    4679   601.4    4875     601    5145   606.6    5317   604.6
#Mann= 3 ,0,0
    1000     .06       0    3583    .035       0    3864     .06       0
#XS Ineff= 5 ,-1
    1000    2220   600.6    2220    3400     610    3400    3583   600.6
    3864    4290     600    4290    5317     610
Permanent Ineff=
       F       F       F       F       F
#Block Obstruct= 2 , 0
                            4099           601.3
Bank Sta=3583,3864
XS Rating Curve= 0 ,0
Exp/Cntr=0.3,0.1

Type RM Length L Ch R = 1 ,38059   ,596.7,640.2,667.6
BEGIN DESCRIPTION:
This cross section corresponds to cross section 38091 of the non-georeferenced CDC model which was the source of this model.
Cross-section modified by USACE February 2007.
Ineffective flow in LOB due to group of structures, effective flow in ROB set at sta 4270.
Old river channel in ROB.
Channel data from 1975 USACE field survey.
END DESCRIPTION:
XS GIS Cut Line= 3
    2299506.1169    6940902.5671   2301072.22401   6938816.13295
   2302044.02292   6937409.74206
#Sta/Elev= 30
    1000   623.5    1038   609.7    1076   611.5    1324   601.9    1484   600.1
    2358   599.4    2385   602.3    2527   597.7    2557   601.7    2636   602.3
    2670   598.7    2718   598.6    2752   601.4    3200   600.5    3417   603.2
    3526   599.2    3640   601.2    3707   579.7 3812.69   571.9    3876   573.8
    3901   579.7    3960   601.4    4449   600.1    4516   583.7    4586   581.2
    4652   581.2    4682   599.3    4807     599    4849   602.8    5319   598.9
#Mann= 3 ,0,0
    1000     .06       0    3640    .035       0    3960     .06       0
#XS Ineff= 5 ,-1
    1000    2360   601.2    2360    3490     610    3490    3640   601.2
    3960    4270   601.4    4270    5319     610
Permanent Ineff=
       F       F       F       F       F
#Block Obstruct= 2 , 0
                            4449           600.1
Bank Sta=3640,3960
XS Rating Curve= 0 ,0
Exp/Cntr=0.3,0.1

Type RM Length L Ch R = 1 ,37419   ,973,982.3,986.1
BEGIN DESCRIPTION:
This cross section corresponds to cross section 37449 of the non-georeferenced CDC model which was the source of this model.
Cross-section modified by USACE February 2007.
Ineffective flow in LOB due to group of structures.
Lockheed Recreation Area in ROB.
Channel data from 1975 USACE field survey.
END DESCRIPTION:
XS GIS Cut Line= 4
   2299506.17596   6940902.58285   2301929.37091   6938851.04594
     2301925.292     6938850.987     2302370.605     6938378.331
#Sta/Elev= 30
    1000   623.5    1005   623.5    1038   609.7    1076   611.7    1327     602
    1405   600.6    1566   599.3    1677   600.1    1805   598.4    1821   599.8
    1876   600.2    2484     600    2496   598.7    2609   600.7    3160   598.7
    3321   599.4    3393   596.7    3527   596.1    3543   598.7    3621   599.4
    3628   599.2    3665   584.1    3734   576.2    3744   573.7 3792.04   570.7
    3863   573.7    3915   584.9    3934   585.9    4004   595.9    4822     598
#Mann= 3 ,0,0
    1000     .06       0    3621    .035       0    4004     .06       0
#XS Ineff= 5 ,-1
    1000    2630   599.4    2630    3440     610    3440    3621   599.4
    4004    4175   595.9    4175    4822     610
Permanent Ineff=
       F       F       F       F       F
Bank Sta=3621,4004
XS Rating Curve= 0 ,0
Exp/Cntr=0.3,0.1

Type RM Length L Ch R = 1 ,36436   ,510,497.7,480
BEGIN DESCRIPTION:
This cross section corresponds to cross section 36466 of the non-georeferenced CDC model which was the source of this model.
Channel data from 1975 USACE field survey.
END DESCRIPTION:
XS GIS Cut Line= 2
   2300102.25187   6941417.19993   2302531.11905   6939651.87898
#Sta/Elev= 30
    1000   614.2    1005   614.2    1041   598.5    1058     598    1078   599.5
    1265   597.4    1840     597    2117     598    2156     597    2172   594.1
    2314   596.8    2700   595.7    2880   597.3    3007   595.6    3208   595.1
    3364   596.5    3486   596.1    3511   587.5    3537   580.4    3591   573.6
 3652.28   570.4    3727   573.6    3748   578.7    3775   589.7    3792     590
    3851   601.9    3891   605.6    3958   608.7    3979   610.7    4003   610.6
#Mann= 3 ,0,0
    1000     .06       0    3486    .035       0    3891     .06       0
Bank Sta=3486,3891
XS Rating Curve= 0 ,0
Exp/Cntr=0.3,0.1

Type RM Length L Ch R = 1 ,35939   ,521,444,385.3
BEGIN DESCRIPTION:
This cross section corresponds to cross section 35969 of the non-georeferenced CDC model which was the source of this model.
Channel data from 1975 USACE field survey.
END DESCRIPTION:
XS GIS Cut Line= 2
    2300693.3081   6941891.10515    2303057.2768   6939777.65334
#Sta/Elev= 30
    1000   611.4    1005   611.4    1028   602.2    1219   601.3    1622   596.8
    1940   595.7    2014   594.4    2079   594.8    2099   591.9    2147   591.7
    2160     594    2339   593.1    2655   595.1    2879     594    3227   594.4
    3246   593.6    3256   590.3    3273     582    3288   577.1    3304   573.6
 3376.18   570.3    3458   573.6    3494   582.9    3515   592.2    3616   597.3
    3828   597.5    3847   600.3    3890   600.4    4083     606    4171   607.3
#Mann= 3 ,0,0
    1000     .06       0    3227    .035       0    3616     .06       0
Bank Sta=3227,3616
XS Rating Curve= 0 ,0
Exp/Cntr=0.3,0.1

Type RM Length L Ch R = 1 ,35495   ,508.6,443,395.8
BEGIN DESCRIPTION:
This cross section corresponds to cross section 35519 of the non-georeferenced CDC model which was the source of this model.
Channel data from 1975 USACE field survey.
END DESCRIPTION:
XS GIS Cut Line= 2
2302071.995496046942383.72166837   2303057.27811   6939777.76423
#Sta/Elev= 30
    1113   596.7    1345     595    1609     595    1719   593.2    1727   594.9
    1764   594.8    1778   593.5    1881   592.5    2197   593.6    2503   592.8
    2566   593.5    2734   590.8    2752   591.5    2770   589.7    2800   591.2
    2854   573.5  2940.3   570.2    3033   573.6    3054   578.7    3091   591.4
    3112   590.6    3139   593.2    3253   592.7    3367   594.8    3598   596.8
    3661   598.2    3701   601.1    3723   601.1    3800   604.9    3899   607.3
#Mann= 3 ,0,0
    1113     .06       0    2800    .035       0    3091     .06       0
Bank Sta=2800,3091
XS Rating Curve= 0 ,0
Exp/Cntr=0.3,0.1

Type RM Length L Ch R = 1 ,35052   ,109.3,118.2,122.7
BEGIN DESCRIPTION:
This cross section corresponds to cross section 35076 of the non-georeferenced CDC model which was the source of this model.
50 feet upstream of channel dam.
Channel data from 1975 USACE field survey.
END DESCRIPTION:
XS GIS Cut Line= 4
2303072.729449086942743.06528603   2303057.34208   6939777.59494
 2303055.4949284 6939421.6380934      2303055.49      6939373.11
#Sta/Elev= 30
    1189     600    1202   599.9    1227   592.9    1270   592.5    1707   593.4
    1728   591.2    1805   590.7    1824   592.6    2314   593.7    2328   594.9
    2746   592.5    2777   590.9    2834   573.5 2936.39   570.1    3042   573.5
    3094     590    3103   590.3    3119   589.1    3133   592.1    3158   592.7
    3408   593.6    3524   595.6    3754   595.4    3922   599.1    3945   601.7
    3960   601.1    3985   603.2    4152   608.8    4546   618.6    4559     620
#Mann= 3 ,0,0
    1189     .06       0    2746    .035       0    3103     .06       0
Bank Sta=2746,3103
XS Rating Curve= 0 ,0
Exp/Cntr=0.3,0.1

Type RM Length L Ch R = 5 ,35000   ,,,
BEGIN DESCRIPTION:
channel dam
crest elevation 573.2
END DESCRIPTION:
Node Name=channel dam
IW Pilot Flow=0
#Inline Weir SE= 2
    2500   573.2    3500   573.2
IW Dist,WD,Coef,Skew,MaxSub,Min_El,Is_Ogee,SpillHt,DesHd
49.5,5,3,0,0.95,, 0 ,,,2,2,
Inline Weir Flap Gates= 0
IW Outlet Rating Curve= 0 ,False,,

Type RM Length L Ch R = 1 ,34934   ,23.9,27.6,29.6
BEGIN DESCRIPTION:
This cross section corresponds to cross section 34957 of the non-georeferenced CDC model which was the source of this model.
43 feet upstream of Bryant-Irvin Road, 55.5 feet downstream of channel dam.
Channel data from 1975 USACE field survey.
END DESCRIPTION:
XS GIS Cut Line= 3
  2303171.707448 6942545.9068369 2303157.7506186  6939856.216303
2303157.012371286939713.94496309
#Sta/Elev= 30
    1421   607.8    1693   595.2    1750   595.1    1792   592.8    1840   593.6
    1871   591.9    1884   593.2    2327   593.9    2347   595.6    2379   595.7
    2411     594    2691   596.4    2720   594.7    2748   589.7    2755   589.8
    2786   577.9    2811   571.2    2828   568.6    2987   568.6    3052   588.8
    3067     592    3092   594.3    3123   592.9    3301   592.1    3377   594.1
    3394   593.1    3826   596.2    3903   597.4    3984   601.2    4253   608.8
#Mann= 3 ,0,0
    1421     .06       0    2691    .035       0    3092     .06       0
#XS Ineff= 2 , 0
            2691   596.4    3092           594.3
Permanent Ineff=
       F       F
Bank Sta=2691,3092
XS Rating Curve= 0 ,0
Exp/Cntr=0.5,0.3

Type RM Length L Ch R = 1 ,34906   ,46.2,49.7,51.9
BEGIN DESCRIPTION:
This cross section corresponds to cross section 34915 of the non-georeferenced CDC model which was the source of this model.
Duplication of previous bridge cross-section without bridge piers.
One-foot upstream of Bryant-Irvin Road.
Bank stations changed by USACE February 2007.
END DESCRIPTION:
XS GIS Cut Line= 5
      2303171.28      6942898.55  2303174.718485 6942779.8316517
     2303186.522     6941229.008     2303187.607     6940864.424
2303208.961237226939482.81133342
#Sta/Elev= 30
    1000   626.9    1146   620.8    1522   598.4    1644     594    1713   592.9
    2014   591.8    2157     593    2243   594.4    2478   601.7 2661.58  603.76
 2661.58   595.8 2683.39   588.2 2691.78     588 2695.97   583.3 2717.95  576.21
 2721.13   571.5    2805   569.9 2895.23  571.38 2898.23  575.89 2929.12     585
 2953.44   596.7 2953.44  603.92    3040   603.3    3252   598.3    3462     595
    3733   596.3    3875   598.3    3997   601.8    4190   609.5    4416   620.1
#Mann= 3 ,0,0
    1000     .06       0 2661.58    .035       0 2953.44     .06       0
Bank Sta=2661.58,2953.44
XS Rating Curve= 0 ,0
Exp/Cntr=0.5,0.3

Type RM Length L Ch R = 3 ,34880   ,,,
BEGIN DESCRIPTION:
Bryant-Irvin Road - south bound
END DESCRIPTION:
Node Name=Bryant-Irvin Roa
Bridge Culvert--1,0,-1,-1, 0
Deck Dist Width WeirC Skew NumUp NumDn MinLoCord MaxHiCord MaxSubmerge Is_Ogee
8.5,35,2.6,0, 14, 14, , , 0.95, 0, 0,0,,
 2661.58 2683.39 2717.95 2720.95 2721.13 2776.66 2779.66    2805 2835.37 2838.37
 2895.23 2898.23 2929.12    2954
  603.76  604.15  604.66  604.71  604.71  605.09  605.11  605.29  605.23  605.22
  604.74  604.71  604.29  603.92
  599.08  599.57  600.08  600.12  600.12  600.47  600.49  600.65   600.6  600.59
  600.13   600.1  599.67  599.18
 2661.58 2683.39 2717.95 2720.95 2721.13 2776.66 2779.66    2805 2835.37 2838.37
 2895.23 2898.23 2929.12    2954
  603.76  604.15  604.66  604.71  604.71  605.09  605.11  605.29  605.23  605.22
  604.74  604.71  604.29  603.92
  599.08  599.57  600.08  600.12  600.12  600.47  600.49  600.65   600.6  600.59
  600.13   600.1  599.67  599.18
Pier Skew, UpSta & Num, DnSta & Num=  ,2719.45, 2 ,2719.45, 2 , 0 , 0 , 0 ,,
       3       3
     560     602
       3       3
     560     602
Pier Skew, UpSta & Num, DnSta & Num=  ,2778.16, 2 ,2778.16, 2 , 0 , 0 , 0 ,,
       3       3
     560     602
       3       3
     560     602
Pier Skew, UpSta & Num, DnSta & Num=  ,2836.87, 2 ,2836.87, 2 , 0 , 0 , 0 ,,
       3       3
     560     602
       3       3
     560     602
Pier Skew, UpSta & Num, DnSta & Num=  ,2896.73, 2 ,2896.73, 2 , 0 , 0 , 0 ,,
       3       3
     560     602
       3       3
     560     602
BR Coef=-1 , 0 , 0 ,1.05, 0 ,,,0.8,-1,0.5,1,
WSPro=,,,, 1 ,,,, 0 ,,,, 0 ,,,,-1 ,-1 ,-1 , 0 , 0 , 0 , 0 , 0
BC Design=,, 0 ,, 0 ,,,,,,
BC HTab HWMax=626.9
BC Use User HTab Curves=0
BC User HTab FreeFlow(D)= 0

Type RM Length L Ch R = 1 ,34856   ,14.3,15.8,17
BEGIN DESCRIPTION:
This cross section corresponds to cross section 34878 of the non-georeferenced CDC model which was the source of this model.
Channel data from 1975 USACE field survey.  Duplication of following bridge cross-section without bridge piers.
Bank stations changed by USACE February 2007.
END DESCRIPTION:
XS GIS Cut Line= 5
      2303204.96      6942894.34  2303207.195843 6942799.2908942
 2303215.5347035 6942403.6342418 2303228.2174235 6941187.5024818
2303241.978059426939478.57568988
#Sta/Elev= 30
    1000   626.9    1146   620.8    1522   598.4    1644     594    1713   592.9
    2014   591.8    2157     593    2243   594.4    2478   601.7 2661.58  603.76
 2661.58   595.8 2683.39   588.2 2691.78     588 2695.97   583.3 2717.95  576.21
 2721.13   571.5    2805   569.9 2895.23  571.38 2898.23  575.89 2929.12     585
 2953.44   596.7 2953.44  603.92    3040   603.3    3252   598.3    3462     595
    3733   596.3    3875   598.3    3997   601.8    4190   609.5    4416   620.1
#Mann= 3 ,0,0
    1000     .06       0 2661.58    .035       0 2953.44     .06       0
#XS Ineff= 2 , 0
         2691.78     588 2929.12             585
Permanent Ineff=
       F       F
Bank Sta=2661.58,2953.44
XS Rating Curve= 0 ,0
Exp/Cntr=0.5,0.3

Type RM Length L Ch R = 1 ,34840   ,46.2,47.9,48.5
BEGIN DESCRIPTION:
This cross section corresponds to cross section 34846 of the non-georeferenced CDC model which was the source of this model.
Duplication of previous bridge cross-section without bridge piers.
One-foot upstream of Bryant-Irvin Road.
Bank stations changed by USACE February 2007.
END DESCRIPTION:
XS GIS Cut Line= 4
2303223.945786546942827.34139884     2303240.198     6941261.185
     2303244.842      6940894.282303256.640458846939388.50133359
#Sta/Elev= 30
    1000   626.9    1125   621.9    1449   602.8    1562   596.9    1661   594.1
    2086   592.2    2239   594.5    2296   595.9    2337     598    2519   602.4
 2581.58   602.1 2581.58   595.8 2601.71   588.3 2617.65   581.4 2635.44  575.58
 2638.44  571.78    2725   569.9 2811.56  571.78 2814.56   574.2 2868.41   595.7
 2868.41  602.06    2940   602.3    3196     599    3305   596.5    3477     595
    3723   595.6    3840   597.1    3958   600.3    4202   609.7    4439     620
#Mann= 3 ,0,0
    1000     .06       0 2581.58    .035       0 2868.41     .06       0
Bank Sta=2581.58,2868.41
XS Rating Curve= 0 ,0
Exp/Cntr=0.5,0.3

Type RM Length L Ch R = 3 ,34824   ,,,
BEGIN DESCRIPTION:
Bryant-Irvin Road - north bound
Downstream bridge: bridge data from 1975 survey.  Minimum low chord elev. 598.3.  Bridge width 30 feet.
Channel data from 1975 USACE field survey.
END DESCRIPTION:
Node Name=Bryant-Irvin Roa
Bridge Culvert--1,0,-1,-1, 0
Deck Dist Width WeirC Skew NumUp NumDn MinLoCord MaxHiCord MaxSubmerge Is_Ogee
3.5,25,2.6,0, 11, 11, , , 0.95, 0, 0,0,,
 2581.58 2635.44 2638.44 2694.14 2697.14    2725 2752.85 2755.85 2811.56 2814.56
    2869
   602.1 602.363 602.378 602.649 602.664   602.8 602.656 602.641 602.353 602.338
  602.06
  598.41 598.391  598.39 598.371  598.37  598.36 598.352 598.351 598.336 598.335
  598.32
 2581.58 2635.44 2638.44 2694.14 2697.14    2725 2752.85 2755.85 2811.56 2814.56
    2869
   602.1 602.363 602.378 602.649 602.664   602.8 602.656 602.641 602.353 602.338
  602.06
  598.41 598.391  598.39 598.371  598.37  598.36 598.352 598.351 598.336 598.335
  598.32
Pier Skew, UpSta & Num, DnSta & Num=  ,2636.94, 2 ,2636.94, 2 , 0 , 0 , 0 ,,
       3       3
     560     600
       3       3
     560     600
Pier Skew, UpSta & Num, DnSta & Num=  ,2695.64, 2 ,2695.64, 2 , 0 , 0 , 0 ,,
       3       3
     560     600
       3       3
     560     600
Pier Skew, UpSta & Num, DnSta & Num=  ,2754.35, 2 ,2754.35, 2 , 0 , 0 , 0 ,,
       3       3
     560     600
       3       3
     560     600
Pier Skew, UpSta & Num, DnSta & Num=  ,2813.06, 2 ,2813.06, 2 , 0 , 0 , 0 ,,
       3       3
     560     600
       3       3
     560     600
BR Coef=-1 , 0 , 0 ,1.05, 0 ,,,0.8,-1,0.5,1,
WSPro=,,,, 1 ,,,, 0 ,,,, 0 ,,,,-1 ,-1 ,-1 , 0 , 0 , 0 , 0 , 0
BC Design=,, 0 ,, 0 ,,,,,,
BC HTab HWMax=626.9
BC Use User HTab Curves=0
BC User HTab FreeFlow(D)= 0

Type RM Length L Ch R = 1 ,34793   ,118.3,114.1,117.2
BEGIN DESCRIPTION:
This cross section corresponds to cross section 34814 of the non-georeferenced CDC model which was the source of this model.
Bridge skewed 33 degrees - bridge area is duplication of
following bridge cross-section without bridge piers.
Channel data from 1975 USACE field survey.
Bank stations changed by USACE February 2007.
END DESCRIPTION:
XS GIS Cut Line= 4
 2303261.09176746942844.41489762 2303269.6729479 6942437.2607985
 2303282.3556679 6941221.12903852303296.974443446939405.63030242
#Sta/Elev= 30
    1000   626.9    1125   621.9    1449   602.8    1562   596.9    1661   594.1
    2086   592.2    2239   594.5    2296   595.9    2337     598    2519   602.4
 2581.58   602.1 2581.58   595.8 2601.71   588.3 2617.65   581.4 2635.44  575.58
 2638.44  571.78    2725   569.9 2811.56  571.78 2814.56   574.2 2868.41   595.7
 2868.41  602.06    2940   602.3    3196     599    3305   596.5    3477     595
    3723   595.6    3840   597.1    3958   600.3    4202   609.7    4439     620
#Mann= 3 ,0,0
    1000     .06       0 2581.58    .035       0 2868.41     .06       0
#XS Ineff= 2 , 0
         2601.71   588.3 2849.12           588.1
Permanent Ineff=
       F       F
Bank Sta=2581.58,2868.41
XS Rating Curve= 0 ,0
Exp/Cntr=0.5,0.3

Type RM Length L Ch R = 1 ,34678   ,547.9,591.3,625.1
BEGIN DESCRIPTION:
This cross section corresponds to cross section 34699 of the non-georeferenced CDC model which was the source of this model.
116 feet downstream of Bryant-Irvin Road.
Effective flow limit in ROB established by USACE October 2006.
Channel data from 1975 USACE field survey.
END DESCRIPTION:
XS GIS Cut Line= 4
   2303356.44713   6942980.68893   2303366.63116   6942497.48386
   2303379.31388    6941281.3521   2303394.54515   6939389.78797
#Sta/Elev= 30
    1000     600    1111     599    1158   595.3    1176   595.6    1207   593.3
    1218     591    1229   585.4    1248   584.5    1286   584.5    1296   591.3
    1328   593.4    1440   595.6    1667     595    1891   596.1    2007   595.6
    2168   592.9    2264     595    2403   595.3    2595   594.7    2665   593.3
    2753   568.5    2774   567.2    2912   567.4    2941   578.6    2991   592.5
    3493   594.8    3858   594.7    4239   603.6    4488   616.4    4591     620
#Mann= 3 ,0,0
    1000     .06       0    2665    .035       0    2991     .06       0
#XS Ineff= 4 ,-1
    1000    1500     600    1500    2665   593.3    2991    3125   592.5
    3125    4591     600
Permanent Ineff=
       F       F       F       F
Bank Sta=2665,2991
XS Rating Curve= 0 ,0
Exp/Cntr=0.3,0.1

Type RM Length L Ch R = 1 ,34087   ,569,535.8,504.8
BEGIN DESCRIPTION:
This cross section corresponds to cross section 34116 of the non-georeferenced CDC model which was the source of this model.
Effective flow limit in ROB established by USACE October 2006.
Drainage channel in LOB removed from conveyance.
Channel data from 1975 USACE field survey.
END DESCRIPTION:
XS GIS Cut Line= 4
   2304047.70198   6943190.78004   2303819.00493   6941714.72295
   2303989.44914   6941065.44013   2303497.05511    6939378.6561
#Sta/Elev= 30
    1000   600.5    1153   596.4    1190   592.3    1238   589.7    1250   582.8
    1277   583.9    1286   589.4    1357   593.3    1443   594.6    1966   594.8
    1996   594.6    2033   592.3    2121   591.3    2353   595.3    2604   595.4
    2634   594.2    2669   580.6    2713   568.2    2736   565.2    2836   565.4
    2874   574.8    2923   592.4    2944   591.6    3043     593    3157     591
    3433     593    4053   593.1    4235     595    4497   599.3    4922     620
#Mann= 3 ,0,0
    1000     .06       0    2604    .035       0    2923     .06       0
#XS Ineff= 3 ,-1
    1000    2604   595.4    2923    3590   592.4    3590    4922     600
Permanent Ineff=
       F       F       F
#Block Obstruct= 2 , 0
            1357   593.3
Bank Sta=2604,2923
XS Rating Curve= 0 ,0
Exp/Cntr=0.3,0.1

Type RM Length L Ch R = 1 ,33551   ,649.6,640.4,635
BEGIN DESCRIPTION:
This cross section corresponds to cross section 33577 of the non-georeferenced CDC model which was the source of this model.
Effective flow limit in ROB established by USACE October 2006.
Drainage channel in LOB removed from conveyance.
Channel data from 1975 USACE field survey.
END DESCRIPTION:
XS GIS Cut Line= 4
    2304766.1779   6943468.66597   2304411.44896   6941883.67997
   2304394.57005   6941000.22012   2303641.18015   6939280.79114
#Sta/Elev= 30
    1000   600.4    1021   599.3    1041   614.9    1063   624.4    1113   625.6
    1374   615.1    1419   599.5    1966   595.2    2025     589    2095   587.7
    2229   593.5    2285   587.9    2298   581.2    2308   580.9    2343     581
    2358   588.7    2404   594.5    2778   594.4    2825   579.7    2862     563
    2990   566.9    3029   574.4    3069   589.2    3250   591.5    3437   589.2
    3552   592.3    4277   591.2    4802   595.5    4936   598.1    5385     620
#Mann= 3 ,0,0
    1000     .06       0    2778    .035       0    3069     .06       0
#XS Ineff= 3 ,-1
    1000    2778   594.4    3069    3980   589.2    3980    5385     600
Permanent Ineff=
       F       F       F
#Block Obstruct= 2 , 0
            2404   594.5
Bank Sta=2778,3069
XS Rating Curve= 0 ,0
Exp/Cntr=0.3,0.1

Type RM Length L Ch R = 1 ,32911   ,127.5,126.4,126.7
BEGIN DESCRIPTION:
This cross section corresponds to cross section 32940 of the non-georeferenced CDC model which was the source of this model.
Cross-section generated from SH 121 Southwest Tollway project study using new topo.  Replaces original cross-section.Effective flow limit in ROB established by USACE October 2006.
---------------------------------------------------------------------
CDC FW111809-01 SH121/SOUTHWEST PARKWAY
CROSS-SECTION 32602 - 32940
UPSTREAM END.
----------------------------------------------
END DESCRIPTION:
XS GIS Cut Line= 3
   2305136.54888   6942700.42111   2305009.22991    6941209.1531
 2304169.8036398 6939379.1891681
#Sta/Elev= 30
    1000     615    1045     612    1060     607    1080     603    1157     601
    1206     600    1725     597    1914     595    1940     594    2010     568
    2019     566    2072     563    2153     563    2180     569    2232     590
    2303     591    2628     591    2700     590    2760     585    2816     583
    2840     585    2950     587    2982     591    3070     591    3200     588
    3289     590    3724     590    4218     594    4428     599    4510     600
#Mann= 3 ,0,0
    1000     .06       0    1940    .035       0    2232     .06       0
#XS Ineff= 3 ,-1
    1000    1940     594    2232    3460     590    3460    4510     600
Permanent Ineff=
       F       F       F
Bank Sta=1940,2232
XS Rating Curve= 0 ,0
Exp/Cntr=0.3,0.1

Type RM Length L Ch R = 1 ,32784   ,21.2,21.4,21.4
BEGIN DESCRIPTION:
This cross section corresponds to cross section 32814 of the non-georeferenced CDC model which was the source of this model.
Interpolated cross-section by USACE 12/1/07.
Paved side slopes of concrete block, natural bottom.
END DESCRIPTION:
XS GIS Cut Line= 3
2305251.616347856942566.71575549       2305132.9      6941189.36
      2304244.23      6939237.33
#Sta/Elev= 30
    1000  614.14 1036.74   612.2 1065.31  609.78 1194.96  603.43 1443.85  599.71
 1714.51  596.73  1767.4  595.73 1834.92  570.01 1863.71     563 1995.93     563
 2000.08  566.62 2017.92  572.13 2060.26  586.55 2078.04  586.55 2098.79  587.41
 2154.12  588.41 2533.51  587.47 2569.07  586.53 2610.57   584.4 2667.87  582.91
 2692.71   583.3 2749.87  585.94 2785.44  590.33 2872.49  590.64 3137.81  589.73
 3252.76     590 3351.56  590.86 4258.68  590.68 4448.22  592.97 4527.26  595.68
#Mann= 6 ,-1,0
    1000     .06       0  1767.4    .018       0 1863.71    .035       0
 1995.93    .018       0 2060.26     .06       0 4527.26     .06       0
Bank Sta=1767.4,2060.26
XS Rating Curve= 0 ,0
Exp/Cntr=0.5,0.3

Type RM Length L Ch R = 1 ,32763   ,192.7,194,193.8
BEGIN DESCRIPTION:
This cross section corresponds to cross section 32794 of the non-georeferenced CDC model which was the source of this model.
Upstream bounding bridge cross-section.
Copy of cross-section 32602 by USACE 12/1/07.  Paved side slopes of concrete block - no change of cross-section template.
Revised Existing Cross Section 32602
USACE relocated 32611 here Dec2006.
END DESCRIPTION:
XS GIS Cut Line= 3
2305271.851324616942559.61834532      2305154.01      6941186.11
      2304253.61      6939232.14
#Sta/Elev= 30
    1000     614    1188     604    1428     600    1689     597    1740     596
    1808     570    1837     563    1971     563    1975     567    2033     586
    2051     586    2072     587    2128     588    2512     587    2548     586
    2590     584    2648   582.7    2694     584    2731     586    2750     589
    2767     591    2964     590    3240     590    3340     591    3700     591
    4065     590    4296     590    4330     591    4450     592    4530     595
#Mann= 5 ,-1,0
    1000     .06       0    1740    .018       0    1837    .035       0
    1971    .018       0    2033     .06       0
#XS Ineff= 2 , 0
            1350  613.43    2344          602.04
Permanent Ineff=
       F       F
Bank Sta=1740,2033
XS Rating Curve= 0 ,0
Exp/Cntr=0.5,0.3

Type RM Length L Ch R = 3 ,32679   ,,,
BEGIN DESCRIPTION:
SH 121/Southwest Parkway
Data from bridge plans.  Concrete block on river side slopes.
END DESCRIPTION:
Node Name=SH 121/SW Parkwa
Bridge Culvert--1,0,-1,-1, 0
Deck Dist Width WeirC Skew NumUp NumDn MinLoCord MaxHiCord MaxSubmerge Is_Ogee
1.5,165,2.6,0, 21, 21, , , 0.95, 0, 0,0,,
    1000    1098    1192    1287    1350    1462    1575    1682 1682.01    1806
    2008    2128 2128.01    2236    2344    2410    2505    2600    3300    4000
    4530
  609.04  609.04  610.41  612.03  613.43  615.76  618.05  619.56  619.56  619.38
  614.98  610.06  610.06  605.99  602.04  599.59  596.62  594.31   592.5   592.3
     592
                                   608.1  610.43     613  614.23     611   612.5
     607     602     605  600.66  596.67
    1000    1098    1192    1287    1350    1462    1575    1682 1682.01    1806
    2008    2128 2128.01    2236    2344    2410    2505    2600    3300    4000
    4530
  609.04  609.04  610.41  612.03  613.43  615.76  618.05  619.56  619.56  619.38
  614.98  610.06  610.06  605.99  602.04  599.59  596.62  594.31   592.5   592.3
     592
                                   608.1  610.43     613  614.23     611   612.5
     607     602     605  600.66  596.67
Pier Skew, UpSta & Num, DnSta & Num=  ,1462, 2 ,1462, 2 , 0 , 0 , 0 ,,
       5       5
     580     620
       5       5
     580     620
Pier Skew, UpSta & Num, DnSta & Num=  ,1570, 2 ,1570, 2 , 0 , 0 , 0 ,,
       5       5
     580     620
      15      15
     580     620
Pier Skew, UpSta & Num, DnSta & Num=  ,1682, 2 ,1682, 2 , 0 , 0 , 0 ,,
       5       5
     580     620
       5       5
     580     620
Pier Skew, UpSta & Num, DnSta & Num=  ,1806, 2 ,1806, 2 , 0 , 0 , 0 ,,
       5       5
     580     620
       5       5
     580     620
Pier Skew, UpSta & Num, DnSta & Num=  ,2008, 2 ,2008, 2 , 0 , 0 , 0 ,,
       5       5
     580     620
       5       5
     580     620
Pier Skew, UpSta & Num, DnSta & Num=  ,2128, 2 ,2128, 2 , 0 , 0 , 0 ,,
       5       5
     580     620
       5       5
     580     620
Pier Skew, UpSta & Num, DnSta & Num=  ,2236, 2 ,2236, 2 , 0 , 0 , 0 ,,
       5       5
     580     620
       5       5
     580     620
BR Coef=-1 , 0 , 0 ,, 0 ,,,0.8,-1,,0,
WSPro=,,,, 1 ,,,, 0 ,,,, 0 ,,,,-1 ,-1 ,-1 , 0 , 0 , 0 , 0 , 0
BC Design=,, 0 ,, 0 ,,,,,,
BC Use User HTab Curves=0
BC User HTab FreeFlow(D)= 0

Type RM Length L Ch R = 1 ,32569   ,223.8,227.1,230.3
BEGIN DESCRIPTION:
This cross section corresponds to cross section 32602 of the non-georeferenced CDC model which was the source of this model.
Downstream bridge bounding cross-section.  Paved side slopes of concrete block - no change of cross-section template. Revised Existing Cross Section 32602.  USACE relocated 32611 here Dec2006.
------------------------------------------------------
CDC FW111809-01 SH121/SOUTHWEST PARKWAY
CROSS-SECTION 32602 - 32940
DOWNSTREAM END.
----------------------------------------------
END DESCRIPTION:
XS GIS Cut Line= 3
2305460.240985066942525.59415373       2305343.7      6941149.03
      2304456.55      6939192.23
#Sta/Elev= 30
    1000     614    1188     604    1428     600    1689     597    1740     596
    1808     570    1837     563    1971     563    1975     567    2033     586
    2051     586    2072     587    2128     588    2512     587    2548     586
    2590     584    2648   582.7    2694     584    2731     586    2750     589
    2767     591    2964     590    3240     590    3340     591    3700     591
    4065     590    4296     590    4330     591    4450     592    4530     595
#Mann= 5 ,-1,0
    1000     .06       0    1740    .018       0    1837    .035       0
    1971    .018       0    2033     .06       0
#XS Ineff= 2 , 0
            1350  613.43    2344          602.04
Permanent Ineff=
       F       F
Bank Sta=1740,2033
XS Rating Curve= 0 ,0
Exp/Cntr=0.5,0.3

Type RM Length L Ch R = 1 ,32342   ,620.9,600.4,585
BEGIN DESCRIPTION:
This cross section corresponds to cross section 32371 of the non-georeferenced CDC model which was the source of this model.
Cross-section generated from SH 121 Southwest Tollway project study using newly topo.  Replaces original cross-section.
Effective flow limit in ROB established by USACE October 2006.
END DESCRIPTION:
XS GIS Cut Line= 3
2305642.604083846942258.56714084   2305567.67204    6940787.4689
      2304490.23      6939183.81
#Sta/Elev= 30
    1000     612    1101     602    1351     599    1461     596    1524     569
    1540     565    1542     563    1681     563    1687     566    1708     569
    1755     588    1773     586    1838     588    1855     585    1875     584
    2074     584    2174     578    2192     578    2238     580    2288     579
    2337     584    2495  586.75    2561     591    2641     594    2672     594
    2765     590    3281     589    4176     590    4301     591    4405     595
#Mann= 3 ,0,0
    1000     .06       0    1461    .035       0    1755     .06       0
#XS Ineff= 3 ,-1
    1000    1461     596    1755    3298     588    3298    4405     600
Permanent Ineff=
       F       F       F
Bank Sta=1461,1755
XS Rating Curve= 0 ,0
Exp/Cntr=0.3,0.1

Type RM Length L Ch R = 1 ,31742   ,877.5,852.6,833.3
BEGIN DESCRIPTION:
This cross section corresponds to cross section 31770 of the non-georeferenced CDC model which was the source of this model.
Effective flow limit in ROB established by USACE October 2006.
Channel data from 1975 USACE field survey.
END DESCRIPTION:
XS GIS Cut Line= 4
   2306266.49216   6941900.40795   2306137.03212   6941282.05092
   2306117.89895   6940089.65009   2306270.41505   6937885.00916
#Sta/Elev= 30
    1000     610    1086     603    1117   602.8    1181   576.5    1220   562.8
 1275.08   558.3    1342   564.4    1366   564.8    1419   579.7    1430   578.7
    1477   581.2    1502   579.9    1542   580.4    1743     588    2373   588.2
    2593   585.8    2777   587.9    3049   588.1    3148   585.1    3200   585.1
    3531   588.2    3930     589    4270   586.1    4557   587.7    4719   586.4
    4849   593.2    4877   599.6    4892   596.8    4941   604.3    5034     610
#Mann= 3 ,0,0
    1000     .06       0    1117    .035       0    1419     .06       0
#XS Ineff= 3 ,-1
    1000    1117   602.8    1419    2775   579.7    2775    5034     600
Permanent Ineff=
       F       F       F
Bank Sta=1117,1419
XS Rating Curve= 0 ,0
Exp/Cntr=0.3,0.1

Type RM Length L Ch R = 1 ,30889   ,680.3,741.2,790.5
BEGIN DESCRIPTION:
This cross section corresponds to cross section 30913 of the non-georeferenced CDC model which was the source of this model.
Effective flow limit in ROB established by USACE October 2006.
Channel data from 1975 USACE field survey.
END DESCRIPTION:
XS GIS Cut Line= 3
   2307042.71207     6941410.571   2306852.94899   6940965.73889
   2306855.10713   6938245.54912
#Sta/Elev= 30
    1000   593.4    1031   592.9    1047   588.2 1112.75   560.7 1186.75   557.3
 1263.75   560.7    1265   562.6    1327     586    1365   587.3    1384   585.6
    1555   586.8    2043   584.9    2376   587.9    2519   586.1    2632   587.7
    2861   585.9    2920   582.8    3042   585.5    3326   584.1    3447   585.2
    3459   583.1    3484     583    3499     585    3617     586    3765   584.1
    3817   585.5    3872   583.8    3904   587.4    4128   590.3    4204     600
#Mann= 3 ,0,0
    1000     .06       0    1031    .035       0    1327     .06       0
#XS Ineff= 3 ,-1
    1000    1031   592.9    1327    1965     586    1965    4204     595
Permanent Ineff=
       F       F       F
Bank Sta=1031,1327
XS Rating Curve= 0 ,0
Exp/Cntr=0.3,0.1

Type RM Length L Ch R = 1 ,30148   ,429.8,514.6,577.8
BEGIN DESCRIPTION:
This cross section corresponds to cross section 30174 of the non-georeferenced CDC model which was the source of this model.
Effective flow limit in ROB established by USACE October 2006.
Channel data from 1975 USACE field survey.
END DESCRIPTION:
XS GIS Cut Line= 3
   2306326.32997   6944087.84911   2307644.36014   6941365.81913
    2307826.3601   6938762.19802
#Sta/Elev= 30
    1000   597.1    1061   593.4    1387   588.4    2086   583.3    2106   585.7
    2486   587.8    2565   583.5    2607   588.1    3777   588.1    4082     587
    4206   582.2    4219   584.2    4267   566.3    4278   565.3 4285.11   559.2
 4357.11   556.4 4432.11   559.2    4436   562.4    4506   587.2    4851     583
    5042   584.9    5121   581.5    5252   585.2    5539   585.5    5856   580.4
    5912   583.1    6155   582.8    6429   586.2    6588   593.8    6634     600
#Mann= 3 ,0,0
    1000     .06       0    4219    .035       0    4506     .06       0
#XS Ineff= 3 ,-1
    1000    4219   584.2    4506    4645   587.2    4645    6634     590
Permanent Ineff=
       F       F       F
Bank Sta=4219,4506
XS Rating Curve= 0 ,0
Exp/Cntr=0.3,0.1

Type RM Length L Ch R = 1 ,29633   ,46.1,45.1,46.1
BEGIN DESCRIPTION:
This cross section corresponds to cross section 29663 of the non-georeferenced CDC model which was the source of this model.
Effective flow limit in ROB established by USACE October 2006.
25 feet upstream of channel dam.
Channel data from 1975 USACE field survey.
END DESCRIPTION:
XS GIS Cut Line= 4
  2306643.936829 6944272.3195512 2308054.4169494 6941285.6073512
 2308724.6117994 6940450.5906412 2309098.2170294 6940164.7906912
#Sta/Elev= 30
    1000     594    1200   589.3    1500   586.2    1800     584    1860   584.1
    2080     582    2120   584.3    2220     586    2560     587    2680     586
    2720     584    2940   584.6    3440   584.3    3860     585    4260     584
    4320     582    4340   573.9    4360   568.1    4380   561.3 4446.79   555.3
 4452.79   555.3    4520   561.7    4540   562.1    4560   570.8    4600     582
    4720     584    5540     584    5620     582    5700     582    5840   590.1
#Mann= 3 ,0,0
    1000     .06       0    4260    .035       0    4720     .06       0
#XS Ineff= 3 ,-1
    1000    4260     584    4720    4725     584    4725    5840     590
Permanent Ineff=
       F       F       F
Bank Sta=4260,4720
XS Rating Curve= 0 ,0
Exp/Cntr=0.3,0.1

Type RM Length L Ch R = 5 ,29625   ,,,
BEGIN DESCRIPTION:
channel dam
crest elevation 561.3
END DESCRIPTION:
Node Name=channel dam
IW Pilot Flow=0
#Inline Weir SE= 2
    4000   561.3    5000   561.3
IW Dist,WD,Coef,Skew,MaxSub,Min_El,Is_Ogee,SpillHt,DesHd
5.5,5,3,0,0.95,, 0 ,,,2,2,
Inline Weir Flap Gates= 0
IW Outlet Rating Curve= 0 ,False,,

Type RM Length L Ch R = 1 ,29588   ,75.5,76.6,79.4
BEGIN DESCRIPTION:
This cross section corresponds to cross section 29613 of the non-georeferenced CDC model which was the source of this model.
Effective flow limit in ROB established by USACE October 2006.
21.5 feet downstream of channel dam.
Channel data from 1975 USACE field survey.
END DESCRIPTION:
XS GIS Cut Line= 4
  2306677.273096 6944302.6838326 2308087.7532162 6941315.9716326
 2308757.9480662 6940480.9549226 2309131.5532962 6940195.1549726
#Sta/Elev= 30
    1000     594    1200   589.3    1500   586.2    1800     584    1860   584.1
    2080     582    2120   584.3    2220     586    2560     587    2680     586
    2720     584    2940   584.6    3860     585    4260     584    4320     582
    4340   573.9    4360   568.1    4380   561.3 4380.51   557.8 4446.51   555.1
 4519.51   557.8    4520   561.7    4540   562.1    4560   570.8    4600     582
    4720     584    5540     584    5620     582    5700     582    5840   590.1
#Mann= 3 ,0,0
    1000     .06       0    4260    .035       0    4720     .06       0
#XS Ineff= 3 ,-1
    1000    4260     584    4720    4725     584    4725    5840     590
Permanent Ineff=
       F       F       F
Bank Sta=4260,4720
XS Rating Curve= 0 ,0
Exp/Cntr=0.3,0.1
