HEC-RAS study CDC_Consolidated_Model.prj: Upper Trinity CDC Consolidated Model

--- CDC_Consolidated_Model.g03 (geometry) --- (continued)

Type RM Length L Ch R = 1 ,218485  ,67,67,67
BEGIN DESCRIPTION:
This cross section corresponds to cross section 218363 of the non-georeferenced CDC model which was the source of this model.
Upstream of Beach Street.
Cross-section generated from points along centrline of Beach Street roadway.
END DESCRIPTION:
XS GIS Cut Line= 6
 2341119.7027942 6961840.9813563 2341119.7027942 6961023.9586464
 2341079.1867654 6960668.8476774 2340676.4099947  6959639.264284
 2340621.5941605 6959424.7678517 2340628.1243955 6957719.9684324
#Sta/Elev= 30
       0  539.77  452.84  533.03  753.35   523.3 1174.86  516.29 1631.55  515.51
 2085.21  510.95 2153.25  511.27 2378.08  517.34 2788.35  526.04 2974.77  525.87
 2984.44     520 3007.66  510.17  3046.8  507.71 3083.02     494 3129.59  484.41
 3282.84  480.16 3310.34  482.75 3336.86     492 3344.51  496.43 3381.33  511.33
 3401.09     512 3444.44  528.62 3589.31     530 3734.17     534 3866.32  539.73
 3990.67     548 4004.26  548.28 4052.54  529.87 4140.35  531.98  4207.5   530.9
#Mann= 4 ,-1,0
       0     .06       0 2378.08    .045       0  3046.8    .035       0
 3381.33     .06       0
#XS Ineff= 2 , 0
       0                 4004.26       0     550
Permanent Ineff=
       F       T
Bank Sta=3046.8,3381.33
XS Rating Curve= 0 ,0
Exp/Cntr=0.5,0.3

Type RM Length L Ch R = 3 ,218450  ,,,
BEGIN DESCRIPTION:
Beach Street
Data from bridge plans, USACE 1975 survey.
Length of bridge 452 feet, minimum low chord elev. 523.  Culvert located at old West Fork oxbow channel not represented due to small size and insignificant impact on flows.
USGS gaging station 08048543 -  Beach Street Gage -   located on downstream side of bridge.  Gage datum elev. 478.70 MSL
END DESCRIPTION:
Node Name=Beach Street
Bridge Culvert--1,0,-1,-1, 0
Deck Dist Width WeirC Skew NumUp NumDn MinLoCord MaxHiCord MaxSubmerge Is_Ogee
1.1,63,2.6,0, 6, 6, , , 0.95, 0, 0,0,,
 2974.77 2974.77 2983.61 3435.61 3435.61 3444.44
     530     530     530     531     531     531
     450     450     523   525.5     450     450
 2974.77 2974.77 2983.61 3435.61 3435.61 3444.44
     530     530     530     531     531     531
     450     450     523   525.5     450     450
Pier Skew, UpSta & Num, DnSta & Num=  ,3036.61, 2 ,3036.61, 2 , 0 , 0 , 0 ,,
       3       3
     450     528
       3       3
     450     528
Pier Skew, UpSta & Num, DnSta & Num=  ,3088.61, 2 ,3088.61, 2 , 0 , 0 , 0 ,,
       3       3
     450     528
       3       3
     450     528
Pier Skew, UpSta & Num, DnSta & Num=  ,3161.61, 2 ,3161.61, 2 , 0 , 0 , 0 ,,
       3       3
     450     528
       3       3
     450     528
Pier Skew, UpSta & Num, DnSta & Num=  ,3251.61, 2 ,3251.61, 2 , 0 , 0 , 0 ,,
       3       3
     450     528
       3       3
     450     528
Pier Skew, UpSta & Num, DnSta & Num=  ,3321.61, 2 ,3321.61, 2 , 0 , 0 , 0 ,,
       3       3
     450     528
       3       3
     450     528
Pier Skew, UpSta & Num, DnSta & Num=  ,3377.61, 2 ,3377.61, 2 , 0 , 0 , 0 ,,
       3       3
     450     528
       3       3
     450     528
BR Coef=-1 , 0 , 0 ,, 0 ,,,0.8,-1,,0,
WSPro=,,,, 1 ,,,, 0 ,,,, 0 ,,,,-1 ,-1 ,-1 , 0 , 0 , 0 , 0 , 0
BC Design=,, 0 ,, 0 ,,,,,,
BC Use User HTab Curves=0
BC User HTab FreeFlow(D)= 0

Type RM Length L Ch R = 1 ,218419  ,47,47,47
BEGIN DESCRIPTION:
This cross section corresponds to cross section 218297 of the non-georeferenced CDC model which was the source of this model.
Downstream of Beach Street.
Cross-section generated from points along centrline of Beach Street roadway.
END DESCRIPTION:
XS GIS Cut Line= 6
 2341180.0614337 6961866.2868327 2341180.0614337 6961049.2641229
  2341139.545405 6960694.1531539 2340736.7686342 6959664.5697604
 2340681.9528001 6959450.0733282  2340688.483035 6957745.2739089
#Sta/Elev= 30
       0  539.77  452.84  533.03  753.35   523.3 1174.86  516.29 1631.55  515.51
 2085.21  510.95 2153.25  511.27 2378.08  517.34 2788.35  526.04 2974.77  525.87
 2984.44     520 3007.66  510.17  3046.8  507.71 3083.02     494 3129.59  484.41
 3282.84  480.16 3310.34  482.75 3336.86     492 3344.51  496.43 3381.33  511.33
 3401.09     512 3444.44  528.62 3589.31     530 3734.17     534 3866.32  539.73
 3990.67     548 4004.26  548.28 4052.54  529.87 4140.35  531.98  4207.5   530.9
#Mann= 4 ,-1,0
       0     .06       0 2378.08    .045       0  3046.8    .035       0
 3381.33     .06       0
#XS Ineff= 2 , 0
       0                 4004.26       0     550
Permanent Ineff=
       F       T
Bank Sta=3046.8,3381.33
XS Rating Curve= 0 ,0
Exp/Cntr=0.5,0.3

Type RM Length L Ch R = 1 ,218372  ,277,277,738
BEGIN DESCRIPTION:
This cross section corresponds to cross section 218250.3 of the non-georeferenced CDC model which was the source of this model.
Ineffective flow in ROB due to Beach Street bridge.
Old West Fork oxbow channel in LOB.
END DESCRIPTION:
XS GIS Cut Line= 6
 2341195.0499155 6961849.8119465 2341178.0685564 6960859.5104318
 2341080.4784064 6960430.1140054 2340924.6108391 6959990.4702451
 2340716.1789835 6959448.9070871   2340731.84128 6957736.5101265
#Sta/Elev= 30
       0  538.58  534.11  529.76  713.89  520.98 1547.19  513.46  1662.9  511.48
 1704.17  505.62 1819.71  500.33 1834.07  502.17 1854.08  514.62 1882.86   512.8
 2271.59  512.41  2433.1  516.31 2737.76  521.43 2892.22  518.23 2964.27     512
 3002.85  507.96 3074.18  485.73 3240.54  479.84 3277.97  485.84 3318.45  499.28
 3340.32   510.8 3414.46  517.75 3473.64  518.28 3709.57  520.38    3780  533.83
 3861.05  539.19 3890.95  535.37  3991.9  536.04 4020.72  531.95 4190.66  531.65
#Mann= 9 ,-1,0
       0     .06       0 1547.19     .08       0 1882.86     .06       0
  2433.1    .045       0 2737.76     .06       0 2964.27    .035       0
 3340.32    .045       0 3473.64     .15       0 3709.57     .04       0
#XS Ineff= 2 ,-1
 1560.34 1854.08     514 3454.52 3861.05     540
Permanent Ineff=
       T       F
Bank Sta=2964.27,3340.32
XS Rating Curve= 0 ,0
Exp/Cntr=0.5,0.3

Type RM Length L Ch R = 1 ,218095  ,252,252,285
BEGIN DESCRIPTION:
This cross section corresponds to cross section 217973.4 of the non-georeferenced CDC model which was the source of this model.
Ineffective flow in ROB due to Beach Street bridge.
Old West Fork oxbow channel in LOB.
END DESCRIPTION:
XS GIS Cut Line= 6
 2341218.3135129 6961837.0169744 2341189.2341134 6960861.1097709
 2340958.6530253 6959981.2964402 2340896.7913874 6959049.5344701
 2341043.3721059 6958699.2899671 2341067.7385303 6957822.2231386
#Sta/Elev= 30
       0  537.86  417.64  532.61  845.23  518.49 1528.41  512.28 1713.74   510.7
 1770.99  503.81 1801.03  493.85  1813.7  493.68 1820.55   488.5 1852.27  490.49
 1862.25  494.86 1884.37  512.32 1892.04  512.52 2514.27  515.55  2828.4  513.87
 2855.96   506.4 2869.07  506.31 2889.04     494 2912.64  487.13 3084.69  480.93
 3103.35  480.94 3126.56  486.55 3168.08  506.23 3181.27  506.36 3192.24  510.55
 3693.07   514.8 3814.69  517.56 3828.32  516.85 3884.65     534 4081.19  536.17
#Mann= 9 ,-1,0
       0     .06       0 1528.41     .15       0 1713.74     .06       0
 1862.25     .15       0 1892.04     .06       0  2828.4    .035       0
 3192.24    .055       0 3693.07     .15       0 3814.69     .04       0
#XS Ineff= 2 ,-1
 3744.83 4081.19     540    1500 1948.62     514
Permanent Ineff=
       F       T
Bank Sta=2828.4,3192.24
XS Rating Curve= 0 ,0
Exp/Cntr=0.3,0.1

Type RM Length L Ch R = 1 ,217842  ,87,87,109
BEGIN DESCRIPTION:
This cross section corresponds to cross section 217720.9 of the non-georeferenced CDC model which was the source of this model.
Upstream of the Beach Street Dam
Ineffective flow in ROB due to Beach Street bridge.
Old West Fork oxbow channel in LOB.
END DESCRIPTION:
XS GIS Cut Line= 4
 2341257.6650071 6961600.1430178 2341126.6147438 6959132.1683299
 2341280.1151285 6958809.9072701 2341298.2227792 6957854.5305144
#Sta/Elev= 30
       0  533.86  188.05  532.16  645.09  519.95 1281.62  512.83  1311.8  508.38
 1427.22   508.1 1467.76  499.21 1589.73  515.35 1691.57  487.29 1710.11     486
 1729.27     486 1765.33  493.02 1791.31   508.3 1811.38  512.94    1817     514
  2467.7  511.12 2524.69  493.54 2541.44  493.67 2576.27  483.98  2633.5  483.42
 2724.94  486.26 2770.29     493 2831.87  509.74 3096.51  509.75 3474.05   516.1
 3589.08  520.34 3649.51  524.59 3670.99  532.35 3695.51  535.52 3783.95  536.92
#Mann= 9 ,-1,0
       0     .06       0 1281.62     .15       0 1589.73     .06       0
 1811.38     .15       0    1817     .06       0  2467.7    .035       0
 2831.87    .055       0 3474.05     .15       0 3589.08     .04       0
#XS Ineff= 3 ,-1
 3701.37 3783.95     540 1589.73    1817     514       0 1589.73  514.89
Permanent Ineff=
       T       T       F
Bank Sta=2467.7,2831.87
XS Rating Curve= 0 ,0
Exp/Cntr=0.3,0.1

Type RM Length L Ch R = 5 ,217764  ,,,
BEGIN DESCRIPTION:
Beach Street Dam
Constructed by TRWD.  Data from TRWD plans.  Top of dam road surface elevation 494.5
-------------------------------
CDC FW112598-01
-------------------------------
END DESCRIPTION:
Node Name=Beach Street Dam
IW Pilot Flow=0
#Inline Weir SE= 2
    2000   494.5    3000   494.5
IW Dist,WD,Coef,Skew,MaxSub,Min_El,Is_Ogee,SpillHt,DesHd
16.55,17.5,3,0,0.95,, 0 ,,,1.5,3,
Inline Weir Flap Gates= 0
IW Outlet Rating Curve= 0 ,False,,

Type RM Length L Ch R = 1 ,217755  ,171,171,175
BEGIN DESCRIPTION:
This cross section corresponds to cross section 217634.1 of the non-georeferenced CDC model which was the source of this model.
Downstream of the Beach Street Dam
Ineffective flow in ROB due to Beach Street bridge.
Old West Fork oxbow channel in LOB.
END DESCRIPTION:
XS GIS Cut Line= 4
 2341294.1528066 6961553.7038469 2341201.1207148  6959175.256239
 2341360.9047637 6958844.0185531 2341378.1774186 6957857.2271061
#Sta/Elev= 30
       0  533.19  913.08  515.52 1215.29  512.54 1312.67  507.07 1399.25  508.72
 1430.41  502.49 1473.62  500.16 1534.78  512.74 1576.34  516.94 1601.05  508.07
 1666.67  498.49 1689.27  485.24 1748.37  492.51 1772.28  513.28  1938.8     514
 2028.56  515.67 2189.08  511.54 2382.91   511.1 2471.61     482 2501.36  479.14
 2583.39  478.91  2647.8     480 2749.55  510.23 2971.46     510 3484.45  517.19
 3555.02  522.17 3606.94  525.21 3634.96     534 3655.21   535.8 3734.97  536.83
#Mann= 8 ,-1,0
       0     .06       0 1576.34     .06       0 1772.28     .15       0
  1938.8     .06       0 2382.91    .035       0 2749.55    .055       0
 3484.45     .15       0 3555.02     .04       0
#XS Ineff= 3 ,-1
 3732.57 3734.97     540       0 1576.34   515.8 1576.34 1772.28  513.28
Permanent Ineff=
       T       F       T
Bank Sta=2382.91,2749.55
XS Rating Curve= 0 ,0
Exp/Cntr=0.3,0.1

Type RM Length L Ch R = 1 ,217585  ,567,567,542
BEGIN DESCRIPTION:
This cross section corresponds to cross section 217463.3 of the non-georeferenced CDC model which was the source of this model.
Old West Fork oxbow channel in LOB.
END DESCRIPTION:
XS GIS Cut Line= 4
 2341314.0552899 6961586.8746092 2341371.7565978 6959232.7533677
 2341501.4763904 6958921.9498088 2341511.3008464 6957859.0822202
#Sta/Elev= 30
       0  532.85 1216.09  509.62 1269.69  504.45 1374.86  504.32  1395.9  499.62
 1425.96  507.07 1515.48   507.6 1577.98  502.96 1618.42  510.17 1676.54  513.33
 1743.66  506.02 1829.43  486.59 1879.61  489.06 1938.12  512.91 1952.73  513.68
 2018.22  515.92 2069.01  511.33 2356.72  511.46 2428.56  484.45 2481.58  479.76
  2610.7     482 2612.62  485.24 2666.89  501.77  2709.9  510.14 3491.71  515.17
 3525.51  512.04  3566.8  522.45 3628.92  527.12 3675.31   535.4 3754.53  536.52
#Mann= 9 ,-1,0
       0     .06       0 1216.09     .15       0 1676.54     .06       0
 1938.12     .15       0 1952.73     .06       0 2356.72    .035       0
  2709.9    .055       0 3491.71     .15       0  3566.8     .04       0
#XS Ineff= 3 ,-1
       0 1676.54  513.33 1676.54    2000  513.33  2709.9 3754.53  510.14
Permanent Ineff=
       F       T       F
Bank Sta=2356.72,2709.9
XS Rating Curve= 0 ,0
Exp/Cntr=0.3,0.1

Type RM Length L Ch R = 1 ,217017  ,1053,1053,1624
BEGIN DESCRIPTION:
This cross section corresponds to cross section 216896 of the non-georeferenced CDC model which was the source of this model.
Located at the old West Fork oxbow channel/modified West Fork river channel confluence.
Effective flow limit set at IH 30 in ROB.
Channel reach length modified to account for reduced effective length for high flows and to better compute volume.
END DESCRIPTION:
XS GIS Cut Line= 4
 2341253.0913925 6961901.0522459 2342019.2238245 6959268.5181783
 2341919.0967963 6958930.0216941 2341980.7879606 6957875.7279476
#Sta/Elev= 30
       0  538.39  239.69  532.74  396.54  532.38 1384.31  510.23  1422.4  509.21
 1449.35     500 1668.52  502.06 1726.75     500 1735.08  503.31 1985.47     502
 2060.22  508.77 2209.14  511.13 2657.96  512.46 2740.98  496.65 2754.44   490.8
 2807.02  484.78 2813.64     480 2838.72  475.07 2906.29  482.41 2996.48     480
 3091.63  509.35 3499.16  509.73 3589.82  508.95  3666.9   498.7 3800.96  507.99
 3865.66  509.02  3926.7  519.05 4024.03  526.52 4087.84  534.89 4150.84  534.67
#Mann= 6 ,-1,0
       0     .06       0 1384.31     .15       0 2657.96     .06       0
 3091.63    .055       0 3499.16     .15       0  3926.7     .04       0
#XS Ineff= 4 ,-1
 4087.84 4150.84     540 3091.63 4087.84  509.35    2325 2657.96  509.35
       0    2325   511.8
Permanent Ineff=
       T       F       F       F
Bank Sta=2657.96,3091.63
XS Rating Curve= 0 ,0
Exp/Cntr=0.3,0.1

Type RM Length L Ch R = 1 ,215964  ,693,693,867
BEGIN DESCRIPTION:
This cross section corresponds to cross section 215842 of the non-georeferenced CDC model which was the source of this model.
Effective flow limit set at IH 30 in ROB.
END DESCRIPTION:
XS GIS Cut Line= 3
 2341170.3212836 6962210.9598793  2342505.236492 6959314.2812891
 2342633.9740205 6957908.2398916
#Sta/Elev= 30
       0  544.07  178.07  539.95   575.7  534.13  613.81  525.87 1507.33  515.28
 1629.06  509.78 1644.08  502.48  1649.3     500 1952.46     500 2025.34  502.21
 2261.55  500.51  2513.1  510.27 2679.11     508 3210.57   509.1 3674.65  510.35
 3876.17  508.22 4030.44  510.22 4038.86  499.16 4057.44     486 4141.53  478.85
  4177.5     482 4214.31  499.49 4233.61  528.22 4237.44     530 4254.42  539.29
 4316.57  545.59 4363.11     551 4413.05  548.93 4467.18  530.98  4601.4  532.26
#Mann= 7 ,-1,0
       0     .09       0  178.07     .06       0 1644.08     .15       0
 3210.57     .06       0 4030.44    .066       0 4237.44     .15       0
 4316.57     .04       0
#XS Ineff= 2 , 0
       0 4030.44   509.7 4363.11       0     551
Permanent Ineff=
       F       T
Bank Sta=4030.44,4237.44
XS Rating Curve= 0 ,0
Exp/Cntr=0.3,0.1

Type RM Length L Ch R = 1 ,215271  ,466,466,741
BEGIN DESCRIPTION:
This cross section corresponds to cross section 215148.4 of the non-georeferenced CDC model which was the source of this model.
END DESCRIPTION:
XS GIS Cut Line= 3
 2341179.0462832 6962330.4915824 2343185.7814011 6959314.2812891
 2343316.6554869 6958014.2659492
#Sta/Elev= 30
       0  545.63  305.62  539.09  364.06  538.31  391.84  531.58  451.61  528.64
  749.37  524.74  758.73  530.51  777.24  531.22  800.72  523.33 1438.23  517.11
 1616.36  510.58 1639.06  503.92 1670.14  502.79 1777.45  505.68  1785.1     500
 1816.35  505.13 1876.16     500 2346.48     500 2354.31  509.24 4326.11  505.31
 4371.08   474.7 4414.87  478.96 4488.89  477.03 4518.69  483.19 4551.33  498.98
 4591.66  510.52 4664.25     514  4787.7   520.6 4834.38     530 4929.37  533.26
#Mann= 5 ,-1,0
       0     .09       0  305.62     .06       0 4326.11    .066       0
 4591.66     .15       0 4664.25     .04       0
#XS Ineff= 2 , 0
       0 4326.11  505.31               0
Permanent Ineff=
       F       F
Bank Sta=4326.11,4591.66
XS Rating Curve= 0 ,0
Exp/Cntr=0.3,0.1

Type RM Length L Ch R = 1 ,214805  ,828,828,1382
BEGIN DESCRIPTION:
This cross section corresponds to cross section 214682.5 of the non-georeferenced CDC model which was the source of this model.
Abandoned sewage treatment plant in LOB - leveed plant blocked for conveyance and storage per CDC Model procedure.
END DESCRIPTION:
XS GIS Cut Line= 3
 2341227.4318329 6962273.2475063 2343527.2944227 6959420.6329964
 2343800.8091512 6958135.2655388
#Sta/Elev= 30
       0  544.48  242.95  539.09  269.56  531.18  402.99  526.86 1394.26  513.77
  1424.5     500 1990.16     500 2008.95  508.87 2101.15  507.15 2116.56     500
 2633.23  508.57  3169.6     506  3356.3   519.2 3616.44     518 3658.13  505.27
 3715.88  517.98 3763.77  505.77 4158.37  512.58 4208.01  506.49 4232.29  492.97
  4318.9  491.46 4406.24  473.22 4490.18  475.09 4519.26  488.71 4531.43  508.06
 4750.39  516.08 4794.87  530.22 4857.87  538.29 4896.91  531.36  4978.4     534
#Mann= 7 ,-1,0
       0     .09       0  242.95     .06       0 3658.13     .04       0
 3715.88      .1       0 4208.01    .066       0 4531.43     .15       0
 4750.39    .035       0
#XS Ineff= 3 ,-1
       0 3298.86  506.49 3709.71 4208.01  506.49 4857.87  4978.4     560
Permanent Ineff=
       F       F       T
#Block Obstruct= 1 ,-1
 3298.86 3709.71     530
Bank Sta=4208.01,4531.43
XS Rating Curve= 0 ,0
Exp/Cntr=0.3,0.1

Type RM Length L Ch R = 1 ,213977  ,1017,1017,2678
BEGIN DESCRIPTION:
This cross section corresponds to cross section 213855 of the non-georeferenced CDC model which was the source of this model.
Abandoned sewage treatment plant in LOB - leveed plant blocked for conveyance and storage per CDC Model procedure.
Channel data estimated from USACE 1975 survey.
END DESCRIPTION:
XS GIS Cut Line= 3
 2341678.0955673 6961796.9975873 2344242.1831846 6959434.2782615
 2344510.6739376 6958440.8620738
#Sta/Elev= 30
       0  522.73   591.8     514   648.3     500 1095.38     500 1104.76   509.7
 1192.13     500 1476.98  509.87 2327.41     506 2448.23  515.62 2488.18  508.91
 2748.65  502.03  2852.1     520 2982.02     520 3155.34  497.86 3232.14  497.86
 3286.71  511.41 3359.31  512.95 3453.01  500.91 3542.15  518.99 3575.82  508.04
 3623.71  506.46 4039.34  512.55 4171.19   507.3 4192.94   484.1 4233.06  482.26
  4246.6   474.3 4296.72  478.48 4321.12  510.83  4459.8  515.54 4515.75  532.41
#Mann= 5 ,-1,0
       0     .06       0 2488.18     .04       0 3542.15      .1       0
 4171.19    .066       0 4321.12    .035       0
#XS Ineff= 2 ,-1
       0 2448.23  507.27 3534.12 4172.55  507.27
Permanent Ineff=
       F       F
#Block Obstruct= 1 ,-1
 2448.23 3534.12     530
Bank Sta=4171.19,4321.12
XS Rating Curve= 0 ,0
Exp/Cntr=0.3,0.1

Type RM Length L Ch R = 1 ,212961  ,495,495,883
BEGIN DESCRIPTION:
This cross section corresponds to cross section 212838.3 of the non-georeferenced CDC model which was the source of this model.
Abandoned sewage treatment plant in LOB - leveed plant blocked for conveyance and storage per CDC Model procedure.
Channel data estimated from USACE 1975 survey.
END DESCRIPTION:
XS GIS Cut Line= 3
 2341481.0248919 6962025.5784969 2345544.3637317 6959071.8156737
 2345653.0846959 6958987.1708755
#Sta/Elev= 30
       0  527.11  779.13  513.93  849.99  511.25  866.52     500  1220.2     500
  1236.5  513.56 1316.04     500 1492.07     500 1565.95  508.74 2458.77  518.02
 2493.41  512.85 3020.44  503.14 3344.24  510.57 3346.61  503.01 3709.93   513.7
 3744.61  519.53 3839.72  515.15 3891.68  504.78 4129.51  507.03 4143.67  514.72
 4179.67  502.36 4246.93  502.39 4250.64  493.22    4290   473.8 4420.25  481.11
 4450.35  504.67 4930.57  512.59 5010.27  519.05  5119.1  551.58 5161.28  554.34
#Mann= 6 ,-1,0
       0     .06       0 2493.41     .04       0 3709.93      .1       0
 4246.93    .066       0 4450.35     .15       0 4930.57    .035       0
#XS Ineff= 2 ,-1
       0 2458.77   507.8 3744.61 4143.67  514.72
Permanent Ineff=
       F       F
#Block Obstruct= 1 ,-1
 2458.77 3744.61     530
Bank Sta=4246.93,4450.35
XS Rating Curve= 0 ,0
Exp/Cntr=0.3,0.1

Type RM Length L Ch R = 1 ,212466  ,1164,1164,1705
BEGIN DESCRIPTION:
This cross section corresponds to cross section 212348.6 of the non-georeferenced CDC model which was the source of this model.
Abandoned sewage treatment plant in LOB - leveed plant blocked for conveyance and storage per CDC Model procedure.
Channel data estimated from USACE 1975 survey.
END DESCRIPTION:
XS GIS Cut Line= 4
 2341561.0009215 6962054.6607484 2343450.1350292 6960790.1569073
 2345826.2791066 6959595.3726873 2346240.3543129 6959393.7880306
#Sta/Elev= 30
       0  525.36  749.14  511.29  818.16     500 1087.04     500 1109.02  512.89
  1182.3     500 1353.86  499.23 1417.98  508.42 2174.81  507.12 2321.34  514.57
 2402.16  506.73 3321.28  509.09 3355.62  508.24 3373.04   519.6 3450.09  501.87
 3948.55  507.13 3998.93  513.72 4040.05  502.77 4099.16  502.78 4122.66  512.31
    4209  509.54 4216.88  487.03  4244.4   473.8  4304.4   473.8 4365.76   486.7
 4503.05   486.8 4550.15  508.26  4785.2     508 5187.22  534.65 5393.43  576.16
#Mann= 5 ,-1,0
       0     .06       0 2321.34     .04       0 3321.28      .1       0
    4209    .066       0 4550.15     .15       0
#XS Ineff= 2 ,-1
       0 2309.83   507.8 3373.04    4209   507.8
Permanent Ineff=
       F       F
#Block Obstruct= 1 ,-1
 2309.83 3373.04     530
Bank Sta=4209,4550.15
XS Rating Curve= 0 ,0
Exp/Cntr=0.3,0.1

Type RM Length L Ch R = 1 ,211302  ,683,683,778
BEGIN DESCRIPTION:
This cross section corresponds to cross section 211182.5 of the non-georeferenced CDC model which was the source of this model.
Abandoned sewage treatment plant in LOB - leveed plant blocked for conveyance and storage per CDC Model procedure.
Channel data estimated from USACE 1975 survey.
END DESCRIPTION:
XS GIS Cut Line= 4
 2341510.1070138 6962163.7187703 2343436.7106666 6961260.0159518
  2346014.283317 6960522.6882172 2346657.4812251 6960381.2802729
#Sta/Elev= 30
       0  528.01    69.1  525.69  617.08  510.82  630.02     500  1040.9     500
 1062.32  510.19 2034.28  508.08 2133.37     512 2152.36  520.43 2175.58  517.05
  2195.8  508.67 3112.83   506.8 3158.62  519.83 3194.44  506.95 3450.14  505.56
 3504.95  494.93 3916.82   496.9 3986.47  499.81 4367.62  498.33 4399.21  505.74
 4811.42  507.85 4841.74  478.14  4852.5   473.5  4922.5   473.5 4987.33  509.01
  5016.5  514.76 5178.91  514.24  5277.4   526.3 5375.34  526.03 5467.54  548.26
#Mann= 10 ,-1,0
       0     .09       0    69.1     .06       0 2175.58     .04       0
 3112.83     .15       0 3504.95      .1       0 3916.82     .15       0
 3986.47      .1       0 4367.62     .15       0 4811.42    .066       0
 4987.33     .15       0
#XS Ineff= 2 ,-1
       0 2152.36  507.85 3158.62 4811.42  507.85
Permanent Ineff=
       F       F
#Block Obstruct= 1 ,-1
 2152.36 3158.62     530
Bank Sta=4811.42,4987.33
XS Rating Curve= 0 ,0
Exp/Cntr=0.3,0.1

Type RM Length L Ch R = 1 ,210619  ,460,460,510
BEGIN DESCRIPTION:
This cross section corresponds to cross section 210502.6 of the non-georeferenced CDC model which was the source of this model.
Channel data estimated from USACE 1975 survey.
Abandoned sewage treatment plant in LOB - leveed plant blocked for conveyance and storage per CDC Model procedure.
END DESCRIPTION:
XS GIS Cut Line= 3
 2341454.8007606 6962220.4300358 2343520.8376922 6961735.8041017
 2347085.7676613 6960984.6257467
#Sta/Elev= 30
       0  530.69  242.43  523.62  571.38     516  684.43     500 1022.18     500
 1047.34  508.97 2591.09     510 2741.27  521.34 2931.66  510.86 3057.89  521.06
 3146.92  505.42 3810.08  506.26 3922.84     494 4157.85     506 4342.17     506
 4426.79     492 4731.47     506 4806.77   500.5 4832.63  481.83  4904.3   473.3
 4953.13  475.66 5006.34  505.19 5059.77   509.8 5069.52  499.51 5166.95  496.72
 5516.78  519.92 5673.95  517.07 5716.91  520.63 5744.46  541.07 5765.34  543.83
#Mann= 6 ,-1,0
       0     .09       0  242.43     .06       0 2741.27     .04       0
 3057.89     .15       0 4806.77    .066       0 5006.34     .15       0
#XS Ineff= 3 ,-1
       0 2445.58     506 3057.89 4752.77     506 5006.34 5765.34  505.19
Permanent Ineff=
       F       F       F
#Block Obstruct= 1 ,-1
 2445.58 3057.89     530
Bank Sta=4806.77,5006.34
XS Rating Curve= 0 ,0
Exp/Cntr=0.3,0.1

Type RM Length L Ch R = 1 ,210160  ,303,303,378
BEGIN DESCRIPTION:
This cross section corresponds to cross section 210038.7 of the non-georeferenced CDC model which was the source of this model.
Channel data estimated from USACE 1975 survey.
END DESCRIPTION:
XS GIS Cut Line= 3
 2341352.7741526 6962454.2407855 2346229.4630691  6961628.956012
 2347035.4406234  6961501.198647
#Sta/Elev= 30
       0  544.99   24.97  544.59   52.05  533.84  101.09     532  667.01  520.96
  862.66  513.45  890.74  501.92 1122.66  502.22 1137.71  507.82 2082.08  506.82
 2264.48  510.27 2853.38     506 3947.32  505.01 4024.75  504.16 4036.74  496.71
 4051.45  496.35 4219.21     498 4380.81  506.18 4477.54  503.94 4561.88     498
 4864.49     506 4939.94  499.23 4948.07  490.04  4999.5   473.1  5039.5   473.1
 5049.88  475.92 5067.43  485.49 5079.05  497.46 5093.82  504.16 5762.07  523.14
#Mann= 5 ,-1,0
       0     .09       0  890.74     .06       0 2853.38     .15       0
 4939.94    .066       0 5093.82     .15       0
#XS Ineff= 2 , 0
       0 4864.49     506               0
Permanent Ineff=
       F       F
Bank Sta=4939.94,5093.82
XS Rating Curve= 0 ,0
Exp/Cntr=0.3,0.1

Type RM Length L Ch R = 1 ,209857  ,628,628,651
BEGIN DESCRIPTION:
This cross section corresponds to cross section 209734 of the non-georeferenced CDC model which was the source of this model.
Channel data estimated from USACE 1975 survey.
END DESCRIPTION:
XS GIS Cut Line= 3
 2341261.9374736 6962626.0030896 2346258.7714086  6961907.385302
 2346859.3999414 6961960.9960956
#Sta/Elev= 30
       0  548.54  112.49  545.73  246.99     534  955.32  515.32  975.59  508.99
 1128.16  499.82 1188.73  504.23    1211  512.45 1829.92  510.16 2979.58  506.23
  3276.8     506 3767.81  505.34 4242.46  504.34 4361.12  496.68 4484.57  503.55
 4506.78  510.44 4574.09     506 4707.55   508.8  4731.6  501.86 4786.92  499.41
 4983.64     504 5046.06  497.71 5051.63  486.28 5071.02  481.54    5157     473
    5177     473 5217.43     508 5359.87  503.65 5592.62  512.42 5651.26  518.94
#Mann= 8 ,-1,0
       0     .09       0 1829.92     .06       0 2979.58     .15       0
  3276.8     .07       0 3767.81     .15       0 5046.06    .066       0
 5217.43     .15       0 5592.62    .035       0
#XS Ineff= 2 , 0
       0  4956.3  504.53 5217.43       0     508
Permanent Ineff=
       F       F
Bank Sta=5046.06,5217.43
XS Rating Curve= 0 ,0
Exp/Cntr=0.3,0.1

Type RM Length L Ch R = 1 ,209229  ,486,486,530
BEGIN DESCRIPTION:
This cross section corresponds to cross section 209098.0 of the non-georeferenced CDC model which was the source of this model.
Channel data estimated from USACE 1975 survey.
END DESCRIPTION:
XS GIS Cut Line= 3
 2341347.3306697 6962978.2497158 2345937.2120771 6962476.5650288
 2346696.4286447 6962430.1366958
#Sta/Elev= 30
       0  545.97  369.96  527.72  973.81  517.38  987.36  509.06 1063.67  500.26
 1097.46  508.75 1164.57  509.78 1465.75  507.76  1969.9  512.49 2156.27  506.62
 2612.57  508.23 3143.47  503.53 3754.96   508.1 3906.85  498.42  3951.7  499.79
 3976.51  507.19 4465.25  504.97 4576.29  510.11 4587.36  493.27  4660.5  485.32
  4685.5  473.19    4697   472.9 4757.99  473.24 4787.19   480.6  4842.9  480.74
 4863.99  494.24 4896.89  498.84 5085.34     498 5141.84  505.98 5377.86     518
#Mann= 8 ,-1,0
       0     .09       0 2156.27     .07       0 2612.57     .15       0
 3143.47     .06       0 3754.96     .15       0 4576.29    .066       0
 4863.99     .15       0 5141.84    .035       0
#XS Ineff= 2 , 0
       0 4576.29     506               0
Permanent Ineff=
       F       F
Bank Sta=4576.29,4863.99
XS Rating Curve= 0 ,0
Exp/Cntr=0.3,0.1

Type RM Length L Ch R = 1 ,208743  ,692,692,173
BEGIN DESCRIPTION:
This cross section corresponds to cross section 208638.1 of the non-georeferenced CDC model which was the source of this model.
Channel data estimated from USACE 1975 survey.
END DESCRIPTION:
XS GIS Cut Line= 3
 2341464.7461685 6963181.0585404 2346581.7108619 6962896.8389868
 2346910.5357426 6962891.7143396
#Sta/Elev= 30
       0   547.9  135.48  536.32  349.21     528   814.6     520  954.12  507.93
 1038.05  509.04 1070.13   513.6 1443.14     514 1619.64  506.21 1807.98  511.59
 2017.54   505.3 2489.48     508  3086.7  503.99 3572.74  502.56 3756.41  506.85
  3833.9  499.19  3984.9  506.47 4564.42  503.16 4572.47  493.24 4595.26  487.17
  4611.3  473.89 4629.93  472.73 4708.56  473.91  4716.2  480.33 4772.24  486.54
 4905.18  487.52 4946.55   504.5 5052.88  503.98 5117.16  511.36 5453.71     524
#Mann= 8 ,-1,0
       0     .09       0 2017.54     .06       0 2489.48     .15       0
  3086.7     .07       0 3756.41     .15       0 4564.42    .072       0
 4946.55     .15       0 5117.16    .035       0
#XS Ineff= 2 , 0
       0 4547.46  505.93               0
Permanent Ineff=
       F       F
Bank Sta=4564.42,4946.55
XS Rating Curve= 0 ,0
Exp/Cntr=0.3,0.1

Type RM Length L Ch R = 1 ,208050  ,1662,1662,6820
BEGIN DESCRIPTION:
This cross section corresponds to cross section 207998 of the non-georeferenced CDC model which was the source of this model.
Channel data estimated from USACE 1975 survey.
Channel reach length modified to account for reduced effective length for high flows and to better compute volume.
END DESCRIPTION:
XS GIS Cut Line= 4
 2341539.4652637 6963415.8896677 2345970.4812343 6963334.7668638
 2346603.8079802 6962936.0056178 2346946.9932305 6962930.3497104
#Sta/Elev= 30
       0  547.16  935.39  512.01  1189.9  514.21 1208.41     508  1243.9  515.38
 1310.05     506 1370.41  516.85 1433.04     504 1928.76  505.22 2507.67  506.84
 2873.18     508 2989.85  498.67 3053.73   504.7 3756.69  505.91 3834.42  498.29
 4086.03  506.38 4111.16  473.65  4145.3  472.53 4279.44  473.62 4285.87  483.08
 4315.92  486.97 4348.92  505.56 4521.96  501.86 4633.87  485.01 4695.14  495.43
 4750.32  483.27 5001.94  501.71 5120.27  501.87 5163.76  511.25  5523.4     524
#Mann= 8 ,-1,0
       0     .09       0 1928.76     .06       0 2507.67     .15       0
 3053.73     .07       0 3756.69     .15       0 4086.03    .072       0
 4348.92     .15       0 5163.76    .035       0
#XS Ineff= 2 , 0
       0 4017.66     506 4348.92       0  505.56
Permanent Ineff=
       F       F
Bank Sta=4086.03,4348.92
XS Rating Curve= 0 ,0
Exp/Cntr=0.5,0.3

Type RM Length L Ch R = 1 ,206389  ,230,230,138
BEGIN DESCRIPTION:
This cross section corresponds to cross section 206448.3 of the non-georeferenced CDC model which was the source of this model.
Upstream of East 1st Street.
Channel data estimated from USACE 1975 survey.
---------------------------------------------------------------------
CDC FW070700-01 Dyer Addition
Located in LOB.
Cross-sections 206448.3 - 209088.06
---------------------------------------------------------------------
END DESCRIPTION:
XS GIS Cut Line= 4
 2341614.8601598  6963472.279432 2345449.1497094 6963553.9425653
 2347221.6992953  6963939.931137 2347885.2533845 6963955.9284139
#Sta/Elev= 30
       0  545.86  495.22  531.49  873.42     514 1122.44  513.09  1132.8  508.03
 1200.06  506.14 1848.69  505.32 2477.39  506.73 2769.83     508 2960.08  498.47
 2976.68  504.66 3724.65   504.2 3864.07  501.21 3915.52  507.65 4150.01  507.27
 4705.57     506 4751.54  501.92 4762.99   482.5    4800     472 4875.04  475.87
 4881.39  481.32  4952.9  504.12 4971.28  501.78 4982.15  498.97 4992.12  507.53
 5066.66  511.82  5590.6  514.62 5609.65  522.14 5861.49   517.8 6312.99  520.59
#Mann= 8 ,-1,0
       0     .09       0 1848.69     .06       0 2477.39     .15       0
 2976.68     .07       0 3724.65     .15       0 4751.54    .066       0
  4952.9     .15       0 4971.28    .035       0
#XS Ineff= 2 , 0
       0                 6312.99       0
Permanent Ineff=
       F       F
Bank Sta=4751.54,4952.9
XS Rating Curve= 0 ,0
Exp/Cntr=0.5,0.3

Type RM Length L Ch R = 3 ,206171  ,,,
BEGIN DESCRIPTION:
East 1st Street
Data from USACE 1975 survey.
Note:  Internal bridge cross-sections modified to represent geometry under bridge.
END DESCRIPTION:
Node Name=East 1st Street
Bridge Culvert--1,0,-1,-1, 0
Deck Dist Width WeirC Skew NumUp NumDn MinLoCord MaxHiCord MaxSubmerge Is_Ogee
110.3,25,2.6,0, 2, 2, , , 0.95, 0, 0,0,,
 4711.04 4914.96
   519.5   519.5
  512.38  512.48
 4711.04 4914.96
   519.5   519.5
  512.38  512.48
Pier Skew, UpSta & Num, DnSta & Num=  ,4772.04, 2 ,4772.04, 2 , 0 , 0 , 0 ,,
       6       6
     450     515
       6       6
     450     515
Pier Skew, UpSta & Num, DnSta & Num=  ,4852.04, 2 ,4852.04, 2 , 0 , 0 , 0 ,,
       6       6
     450     515
       6       6
     450     515
BR Coef=-1 , 0 , 0 ,, 0 ,,,0.8,-1,,0,
WSPro=,,,, 1 ,,,, 0 ,,,, 0 ,,,,-1 ,-1 ,-1 , 0 , 0 , 0 , 0 , 0
BR U #Sta/Elev= 492
       0  548.23     .68  548.22   26.63   547.6   27.12   547.6   52.94  546.99
   53.64  546.98   80.06  546.35  105.64  545.75  162.76     544  171.86  543.86
  211.57  542.72  231.62     542  238.86  541.94  254.87  541.48  270.84  541.01
  301.83  540.12  348.43  538.63  360.89  538.22   364.2  538.08  364.98   538.1
  393.81  537.18  396.27  537.09  401.23  537.12  401.85  536.89   423.5  536.11
  426.57  535.99  471.45  534.37  478.54  534.06  480.08  534.02  521.09   532.3
  526.97  531.96  530.23  531.92   542.2  531.41  543.35  531.34  571.34  530.16
  574.93  529.98  588.42  529.39  600.27  528.86  611.35  528.39  619.77  528.05
  625.98  527.69  629.29  527.53  653.23  526.46  659.35  526.18  662.23     526
  675.29  525.33  676.51  525.35  696.28  524.38  708.11  523.81  713.31  523.51
   718.9  523.28  729.93  522.75  744.06     522  759.93  521.24  766.58  520.91
   767.2  520.93  775.99  520.49  784.52     520  817.55  518.52  821.63  518.31
  873.18  516.03  875.77  515.95  880.24  515.73  880.66  515.66  887.62  515.32
  894.53  514.96  894.88  515.05  907.57  514.48  911.05  514.48  913.81  514.38
  944.92  513.38   975.2  512.43  983.79  512.15  992.43  511.97  996.47  511.75
 1008.81  511.36    1014  511.31 1056.69  509.98 1059.18  510.13  1072.4     510
  1080.1  509.75  1106.4  509.28  1119.5  509.04 1123.71  509.41 1125.76  509.94
 1127.82  509.32 1132.46  508.04 1134.21     508 1135.66  507.66  1142.1  507.51
 1145.23  507.48 1157.49  507.47 1181.85  506.99 1194.92  506.98 1222.42  506.45
 1236.26  506.44  1248.7  506.35 1252.43  506.08 1259.65   505.9 1267.88  505.89
 1271.51   505.6 1277.21  505.72  1286.3  505.66 1291.02  505.68 1292.98  505.64
 1298.38  505.61 1302.78  505.51 1308.31  505.48 1312.57  505.39 1318.34  505.36
 1322.47  505.28 1336.45   505.2 1350.87   505.1 1364.84  505.02 1365.34  504.99
 1372.72  504.95 1406.64  504.74 1420.29  504.64 1438.49  504.56  1467.8  504.46
 1483.46  504.38 1507.54  504.38 1518.44   504.4  1529.6   504.4 1540.82  504.42
 1566.07  504.43 1577.53  504.45  1598.2  504.45 1599.99  504.46 1618.06  504.46
 1644.37  504.48 1664.86  504.48 1686.21   504.5 1702.13   504.5 1703.67  504.51
 1721.45  504.51 1729.55  504.52 1750.18  504.69 1769.61  504.84 1816.08  505.23
 1826.01   505.3 1835.91  505.39  1869.8  505.66 1890.25  505.83 1899.43  505.89
 1911.13  506.03  1921.1  506.08 1925.48  506.07 1928.99     506 1937.39  506.07
 1937.53  506.44 1963.88   506.8 1971.65   506.9 2017.44  506.92 2043.85  506.94
 2054.01  506.94 2117.31  506.98  2143.9  507.02 2170.31  507.07 2187.23  507.09
 2194.71  507.11 2218.62  507.15 2236.69  507.15 2238.36  507.16 2256.36  507.16
 2258.73  507.17 2277.34  507.17 2284.32  507.18 2312.38  507.18 2313.98  507.19
 2334.23  507.19 2387.86  507.25 2396.26  507.25 2407.53  507.27 2416.05  507.27
 2446.08  507.31 2453.59  507.31 2478.63  507.35 2488.36  507.44 2493.46  507.46
 2511.34  507.62 2517.63  507.66 2522.86  507.72 2544.98   507.9 2557.96  507.97
 2568.12  507.99 2598.98     508 2609.65  508.01  2628.1  508.01 2676.41  508.04
 2706.41  508.05 2726.55  508.07 2745.67  508.08 2752.97  508.11 2770.37  508.13
 2779.42  508.15 2785.39  507.98 2789.73  507.97  2812.7  508.02 2827.69  508.06
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BR U #Mann= 3
       0     .06 4711.04    .055 4914.96     .06
BR U Banks=4711.04,4914.96
BR D #Sta/Elev= 492
       0  548.23     .68  548.22   26.63   547.6   27.12   547.6   52.94  546.99
   53.64  546.98   80.06  546.35  105.64  545.75  162.76     544  171.86  543.86
  211.57  542.72  231.62     542  238.86  541.94  254.87  541.48  270.84  541.01
  301.83  540.12  348.43  538.63  360.89  538.22   364.2  538.08  364.98   538.1
  393.81  537.18  396.27  537.09  401.23  537.12  401.85  536.89   423.5  536.11
  426.57  535.99  471.45  534.37  478.54  534.06  480.08  534.02  521.09   532.3
  526.97  531.96  530.23  531.92   542.2  531.41  543.35  531.34  571.34  530.16
  574.93  529.98  588.42  529.39  600.27  528.86  611.35  528.39  619.77  528.05
  625.98  527.69  629.29  527.53  653.23  526.46  659.35  526.18  662.23     526
  675.29  525.33  676.51  525.35  696.28  524.38  708.11  523.81  713.31  523.51
   718.9  523.28  729.93  522.75  744.06     522  759.93  521.24  766.58  520.91
   767.2  520.93  775.99  520.49  784.52     520  817.55  518.52  821.63  518.31
  873.18  516.03  875.77  515.95  880.24  515.73  880.66  515.66  887.62  515.32
  894.53  514.96  894.88  515.05  907.57  514.48  911.05  514.48  913.81  514.38
  944.92  513.38   975.2  512.43  983.79  512.15  992.43  511.97  996.47  511.75
 1008.81  511.36    1014  511.31 1056.69  509.98 1059.18  510.13  1072.4     510
  1080.1  509.75  1106.4  509.28  1119.5  509.04 1123.71  509.41 1125.76  509.94
 1127.82  509.32 1132.46  508.04 1134.21     508 1135.66  507.66  1142.1  507.51
 1145.23  507.48 1157.49  507.47 1181.85  506.99 1194.92  506.98 1222.42  506.45
 1236.26  506.44  1248.7  506.35 1252.43  506.08 1259.65   505.9 1267.88  505.89
 1271.51   505.6 1277.21  505.72  1286.3  505.66 1291.02  505.68 1292.98  505.64
 1298.38  505.61 1302.78  505.51 1308.31  505.48 1312.57  505.39 1318.34  505.36
 1322.47  505.28 1336.45   505.2 1350.87   505.1 1364.84  505.02 1365.34  504.99
 1372.72  504.95 1406.64  504.74 1420.29  504.64 1438.49  504.56  1467.8  504.46
 1483.46  504.38 1507.54  504.38 1518.44   504.4  1529.6   504.4 1540.82  504.42
 1566.07  504.43 1577.53  504.45  1598.2  504.45 1599.99  504.46 1618.06  504.46
 1644.37  504.48 1664.86  504.48 1686.21   504.5 1702.13   504.5 1703.67  504.51
 1721.45  504.51 1729.55  504.52 1750.18  504.69 1769.61  504.84 1816.08  505.23
 1826.01   505.3 1835.91  505.39  1869.8  505.66 1890.25  505.83 1899.43  505.89
 1911.13  506.03  1921.1  506.08 1925.48  506.07 1928.99     506 1937.39  506.07
 1937.53  506.44 1963.88   506.8 1971.65   506.9 2017.44  506.92 2043.85  506.94
 2054.01  506.94 2117.31  506.98  2143.9  507.02 2170.31  507.07 2187.23  507.09
 2194.71  507.11 2218.62  507.15 2236.69  507.15 2238.36  507.16 2256.36  507.16
 2258.73  507.17 2277.34  507.17 2284.32  507.18 2312.38  507.18 2313.98  507.19
 2334.23  507.19 2387.86  507.25 2396.26  507.25 2407.53  507.27 2416.05  507.27
 2446.08  507.31 2453.59  507.31 2478.63  507.35 2488.36  507.44 2493.46  507.46
 2511.34  507.62 2517.63  507.66 2522.86  507.72 2544.98   507.9 2557.96  507.97
 2568.12  507.99 2598.98     508 2609.65  508.01  2628.1  508.01 2676.41  508.04
 2706.41  508.05 2726.55  508.07 2745.67  508.08 2752.97  508.11 2770.37  508.13
 2779.42  508.15 2785.39  507.98 2789.73  507.97  2812.7  508.02 2827.69  508.06
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BR D #Mann= 3
       0     .06 4711.04    .055 4914.96     .06
BR D Banks=4711.04,4914.96
BC Design=,, 0 ,, 0 ,,,,,,
BC Use User HTab Curves=0
BC User HTab FreeFlow(D)= 0

Type RM Length L Ch R = 1 ,206158  ,0,0,0
BEGIN DESCRIPTION:
This cross section corresponds to cross section 206218.0 of the non-georeferenced CDC model which was the source of this model.
Downstream of East 1st Street.
Central City model begins here.
********************************************** Rating curve as downstream condition developed from the current Upper Trinity River CDC Model.
**********************************************
Channel data estimated from USACE 1975 survey.
END DESCRIPTION:
XS GIS Cut Line= 6
     2341904.096     6963632.544     2343430.684     6963683.607
     2344852.789     6963698.881     2345465.415      6963790.52
     2347058.227     6964146.116     2347947.115     6964085.101
#Sta/Elev= 30
       0  546.85  369.23   548.9  512.04  541.71  562.18  536.03  572.53  544.23
  603.81  533.98  663.08  540.28  684.12  537.77  686.41     530  788.51  524.26
  821.63  512.25 1096.67     506  1177.8   497.8 1490.48   497.8  1532.1  504.55
 2227.97  504.14 2413.28  504.51 2932.16  493.48 3128.06  502.57 3345.99  497.58
 3560.99  505.16 4383.29     506 4429.29  502.89 4488.22  473.47 4503.96     472
 4559.71  473.37 4635.51  509.09 4886.06  506.87 4979.55  513.78 6093.63     520
#Mann= 7 ,-1,0
       0     .09       0  512.04     .15       0 2227.97     .06       0
 2413.28     .15       0 4383.29    .066       0 4635.51     .15       0
 4979.55    .035       0
#XS Ineff= 2 , 0
       0                 6093.63       0
Permanent Ineff=
       F       F
Bank Sta=4383.29,4635.51
XS Rating Curve= 0 ,0
Exp/Cntr=0.5,0.3
Stream Node=Clear Fork      ,cf              , 0 , 0 ,Upstream end
Stream Node=Clear Fork      ,cf              , 0 , 1 ,Downstream end
Stream Node=West Fork       ,wf4             , 0 , 0 ,Upstream end
Stream Node=West Fork       ,wf4             , 0 , 1 ,Downstream end
Stream Node=West Fork       ,wf3             , 0 , 0 ,Upstream end
Stream Node=West Fork       ,wf3             , 0 , 1 ,Downstream end
LCMann Table=0

--- CDC_Consolidated_Model.g04 (geometry) ---

Geom Title=Exist: 1%+ AEP [WF/EF/TRMS]
Program Version=6.60
BEGIN GEOM DESCRIPTION:
Existing: Geometry file for use with 1%+ AEP peak flows for the WF/EF/TRMS
END GEOM DESCRIPTION:

Junct Name=ef-wf
Junct Desc=, 0 , 0 , 0 ,0
Up River,Reach=Elm Fork        ,ef3 ds
Up River,Reach=West Fork       ,wf
Dn River,Reach=Main Stem       ,ms
Junc L&A=3030,20
Junc L&A=1494,0

Junct Name=J2
Junct Desc=, 0 , 0 ,-1 ,0
Up River,Reach=Elm Fork        ,ef3
Dn River,Reach=Elm Fork        ,PGBT split west
Dn River,Reach=Elm Fork        ,PGBT split east
Junc L&A=741,0
Junc L&A=370,0

Junct Name=J1
Junct Desc=, 0 , 0 ,-1 ,0
Up River,Reach=Elm Fork        ,PGBT split west
Up River,Reach=Elm Fork        ,PGBT split east
Dn River,Reach=Elm Fork        ,ef3 ds
Junc L&A=1067,0
Junc L&A=1067,0

River Reach=Elm Fork        ,ef3
Reach XY= 30
      2443507.86      7054781.77      2443915.37      7053909.89
      2443712.82      7053314.17      2443133.27      7052713.75
      2443336.18      7052124.19       2443690.1      7052046.36
      2444983.67      7052568.29      2445822.43      7052571.42
      2446558.92      7052244.63      2446983.77      7051618.15
      2446833.53      7051182.86      2445539.52      7051137.95
      2445258.66      7050815.85      2446648.28      7050138.14
      2446851.94      7049721.91      2446747.18      7049390.79
      2445718.34      7049007.95      2445520.89      7048288.45
      2444349.09      7048317.26      2443701.18      7047191.54
      2443845.71      7046976.55      2446154.44      7046114.48
      2446441.34      7045466.69      2446602.22      7043949.82
      2448092.76      7043729.22      2448101.07      7043184.86
      2447026.42      7042543.32      2447988.56      7041959.85
      2447709.25      7040463.12      2447850.52      7040050.17

Type RM Length L Ch R = 1 ,107977  ,37,107,201
BEGIN DESCRIPTION:
This cross section corresponds to cross section 107964 of the non-georeferenced CDC model which was the source of this model.
FIS SECTION RECODED BY OEI, Added dense shrubs b/w fairways, mounds b/s 6 & 8
END DESCRIPTION:
XS GIS Cut Line= 6
2445808.357103357046657.124288962445775.275148517046645.97208031
2445068.484895417046738.446960972444833.605115837046686.63210396
2442716.03290743 7046775.21001082441539.11334527 7046806.0485318
#Sta/Elev= 30
    1015     454    1065   437.6    1395     438    1465     444    1600     448
  1819.3     446    1880     436    1903   424.7    1925  422.71    1943  422.71
  1951.5     436  1972.4     442    2100     446    2185     446    2215     450
    2515     446    2575     447    2610     451    2640     446    3033     445
    3072     439    3109     446    3280   446.2    3381     444    3444     446
    3775     446    3859     447    3905     444    5215     444    5300     458
#Mann= 12 ,-1,0
    1015     .04       0    1395     .12       0  1819.3     .05       0
    2100     .12       0    2640     .05       0    3033     .09       0
    3109     .12       0    3280     .05       0    3444     .12       0
    3775     .05       0    3859      .1       0    3905     .06       0
#XS Ineff= 2 ,-1
    1015  1819.3     446    2100    5300     446
Permanent Ineff=
       F       F
#Block Obstruct= 1 ,-1
    3033    3109     442
Bank Sta=1819.3,2100
XS Rating Curve= 0 ,0
Exp/Cntr=0.3,0.1

Type RM Length L Ch R = 1 ,107870  ,759,1177,557
BEGIN DESCRIPTION:
This cross section corresponds to cross section 107820 of the non-georeferenced CDC model which was the source of this model.
NEW SECTION ADDED BY OEI
----------------------------------------
CDC LEW050102-01 Vista Ridge Golf Center
Cross-section 107820 - 109670
Located in ROB.
----------------------------------------
END DESCRIPTION:
XS GIS Cut Line= 6
2446120.972947937046749.88591446 2445827.42858757046622.02593397
2445390.500983697046619.73591229 2445120.92442317046650.20566763
2444876.301224687046604.346507392441393.439424017046715.47030088
#Sta/Elev= 30
       0     460     145     440     190     438     770   437.6     820     446
     860     448    1055     446    1069     440    1102     436    1140  422.43
    1158  422.43    1209     442    1240   445.3    1325     444    1660     442
    1810     446    2015     446    2066     437    2105     447    2165     451
    2190     447    2230     447    2242     450    2288     446    2460     446
    2520     446    2526     442    2900     444    4640     444    4762     452
#Mann= 9 ,-1,0
       0     .04       0     770     .12       0    1055     .05       0
    1240     .05       0    1325      .1       0    2015     .09       0
    2105     .05       0    2460      .1       0    2900     .06       0
#XS Ineff= 2 ,-1
     120    1060     446    1240    4762   445.3
Permanent Ineff=
       F       F
#Block Obstruct= 1 ,-1
    2015    2105     442
Bank Sta=1055,1240
XS Rating Curve= 0 ,0
Exp/Cntr=0.3,0.1

Type RM Length L Ch R = 1 ,106693  ,24,24,24
BEGIN DESCRIPTION:
This cross section corresponds to cross section 106700 of the non-georeferenced CDC model which was the source of this model.
Water tank section DS Copied section
END DESCRIPTION:
XS GIS Cut Line= 5
2446254.662969267046465.101050972445876.386822917045960.52594464
2445562.02557501 7045963.65257882445240.248987597045964.12501881
2440747.161517087045998.48026505
#Sta/Elev= 30
     990     458     990     444    1003   439.7    1038   436.3    1169   436.2
    1193   440.7    1241     441    1279   424.7    1300   420.2    1317   420.2
    1336   433.2    1360   439.5    1390   441.6    1417   446.9    1489   447.7
    2142   446.1    2438     448    2882     446    3022   448.6    4190   446.7
    4252   443.9    4269   446.4    5068   445.2    5380   442.3    6015     446
    6133   450.6    6161   445.7    6716   447.6    6737   447.9    6750     458
#Mann= 4 ,-1,0
     990     .06       0    1241     .05       0    1390     .12       0
    2142     .06       0
#XS Ineff= 3 ,-1
     200    1241     441    1390    1500   441.6    6133    6750     451
Permanent Ineff=
       F       F       F
#Block Obstruct= 1 ,-1
    6165    6665     453
Bank Sta=1241,1390
XS Rating Curve= 0 ,0
Exp/Cntr=0.3,0.1

Type RM Length L Ch R = 1 ,106669  ,850,721,560
BEGIN DESCRIPTION:
This cross section corresponds to cross section 106657 of the non-georeferenced CDC model which was the source of this model.
Water tank section DS
-------------------------------------------------
CDC LEW052401-1 Water Storage Tank
Cross-section 106657 - 107964
Project located in far ROB west of Gun Club road.
-------------------------------------------------
END DESCRIPTION:
XS GIS Cut Line= 3
2446264.197070937046450.406198472445896.118082677045935.09522122
2440769.508913347045970.63287979
#Sta/Elev= 30
     990     458     990     444    1003   439.7    1038   436.3    1169   436.2
    1193   440.7    1241     441    1279   424.7    1300   420.2    1317   420.2
    1336   433.2    1360   439.5    1390   441.6    1417   446.9    1489   447.7
    2142   446.1    2438     448    2882     446    3022   448.6    4190   446.7
    4252   443.9    4269   446.4    5068   445.2    5380   442.3    6015     446
    6133   450.6    6161   445.7    6716   447.6    6737   447.9    6750     458
#Mann= 4 ,-1,0
     990     .06       0    1241     .05       0    1390     .12       0
    2142     .06       0
#XS Ineff= 3 ,-1
     200    1241     441    1390    1500   441.6    6133    6750     451
Permanent Ineff=
       F       F       F
Bank Sta=1241,1390
XS Rating Curve= 0 ,0
Exp/Cntr=0.3,0.1
