HEC-RAS study CDC_Consolidated_Model.prj: Upper Trinity CDC Consolidated Model

--- CDC_Consolidated_Model.g13 (geometry) --- (continued)

Type RM Length L Ch R = 1 ,40693   ,12,63,68
XS GIS Cut Line= 3
  2435290.1016926975511.634309312434474.129470716967013.45722598
2434545.093012366962463.18234172
#Sta/Elev= 30
    1670  439.93 1812.14     433 2169.54  434.69 2212.32     426 2234.17     432
 2653.03     433 2676.98  427.12 2700.92  432.67 2760.47     426 2770.82     433
 3353.06  430.94 3569.02  422.94  3833.7  429.99  5499.9     426 5551.96  439.94
 5691.47  437.94 5746.19     44910012.77     44810084.28     43210349.98  414.79
10650.77     41510891.76     43311348.09  428.0111703.63     43411851.56  404.57
11901.48  409.6911938.51     43412241.42     43612310.07  444.4812419.88  448.25
#Mann= 13 ,-1,0
    1670    .065       0 2234.17     .08       0 2700.92     .05       0
 2770.82    .075       0 3353.06     .04       0  3833.7    .075       0
10012.77    .035       010084.28    .045       010891.76    .085       0
11703.63     .05       011938.51     .08       012241.42     .05       0
12310.07     .08       0
#XS Ineff= 2 , 0
        11662.18     435
Permanent Ineff=
       F       F
Bank Sta=11703.63,11938.51
XS Rating Curve= 0 ,0
Exp/Cntr=0.3,0.1

Type RM Length L Ch R = 1 ,40633   ,22,112,121
XS GIS Cut Line= 3
  2435299.6123266975510.40998928 2434487.98038226967027.33707263
2434606.614641466962485.95975782
#Sta/Elev= 30
    1694  439.95 2290.53     427 2395.95     432 2632.35     433 2648.66     426
 2742.57     433 3377.01  430.94 3592.74  422.94 3859.34  430.07 5509.98  424.94
 5560.07  439.94 5701.11  437.94 5757.96     44910019.74     44810113.91     430
10370.41     41410645.94     41510889.97     43311706.15     43411754.64     429
11795.54  409.6611857.06  404.5811911.57     40911929.25     430 11953.3     434
12022.33     42412206.95     42412253.15  435.6312355.36  443.9912426.37  448.16
#Mann= 13 ,-1,0
    1694    .065       0 2395.95     .08       0 2632.35     .05       0
 2742.57    .075       0 3377.01     .04       0 3859.34    .075       0
10019.74    .035       010113.91    .045       010889.97    .085       0
11706.15     .05       0 11953.3     .09       012253.15     .05       0
12355.36     .08       0
#XS Ineff= 2 , 0
        11706.15     434
Permanent Ineff=
       F       F
Bank Sta=11706.15,11953.3
XS Rating Curve= 0 ,0
Exp/Cntr=0.3,0.1

Type RM Length L Ch R = 1 ,40527   ,17,87,95
XS GIS Cut Line= 3
  2435305.9780676975508.74621613 2434497.9485535 6967027.7566328
2434692.197685456962502.40941058
#Sta/Elev= 30
    1733  439.21 2341.23     427 2472.76     432 2634.27     433  2643.9     426
 2749.81     433 3394.86     431  3611.5  422.94 3925.91  430.62 5504.33  424.94
 5562.12  438.94 5708.17  437.94 5767.98   447.410029.35  447.0510117.64     430
10351.24  415.0210686.23  414.21 10896.6  432.5211727.33     43411760.09     433
11802.28     41211855.18   404.6 11906.3     410 11921.7     42511964.08     434
12014.43     42412205.89     42412246.95  435.26 12357.8     444 12429.6     448
#Mann= 13 ,-1,0
    1733    .065       0 2472.76     .08       0 2634.27     .05       0
 2749.81    .075       0 3394.86     .04       0 3925.91    .075       0
10029.35    .035       010117.64    .045       0 10896.6    .085       0
11727.33     .05       011964.08     .09       012246.95     .05       0
 12357.8     .08       0
#XS Ineff= 2 , 0
        11727.33     434
Permanent Ineff=
       F       F
Bank Sta=11727.33,11964.08
XS Rating Curve= 0 ,0
Exp/Cntr=0.3,0.1

Type RM Length L Ch R = 1 ,40444   ,17,85,93
XS GIS Cut Line= 3
  2435311.0778936975507.791355012434506.954629876967032.68284808
2434784.168171556962518.86629717
#Sta/Elev= 30
    1760  438.58 2379.78     427 2533.23     432 2672.55     433 2679.13     426
 2724.43     433  2749.6     426 3410.55  430.94 3679.79  422.94 3908.19     431
 5504.36  424.94 5562.23  438.94 5700.55  436.94 5760.25     44810026.44     448
10092.04     43210198.42     42010459.55  414.0110723.36     41510888.56     433
11772.99     43411807.51  408.6611845.23  404.6211919.78  412.3811961.77  431.08
12127.82     42412251.74  434.4512285.92     44312343.43     44412441.25     448
#Mann= 13 ,-1,0
    1760    .065       0 2533.23     .08       0 2672.55     .05       0
 2724.43    .075       0 3410.55     .04       0 3908.19    .075       0
10026.44    .035       010092.04    .045       010888.56    .085       0
11772.99     .05       011961.77     .09       012251.74     .05       0
12343.43     .08       0
#XS Ineff= 2 , 0
        11772.99     434
Permanent Ineff=
       F       F
Bank Sta=11772.99,11961.77
XS Rating Curve= 0 ,0
Exp/Cntr=0.3,0.1

Type RM Length L Ch R = 1 ,40362   ,19,100,108
BEGIN DESCRIPTION:
---------------------------------------------------------------------
CDC GP072315-1 IH-30 Westbound Frontage Road
Cross-sections 40362 - 40693.  Mitigation swale in ROB.
---------------------------------------------------------------------
END DESCRIPTION:
XS GIS Cut Line= 3
  2435316.358565 6975506.51097312434514.231828996967034.24534805
2434874.516840526962527.95049849
#Sta/Elev= 30
    1770  437.77 2497.34     427 2623.55     433 2738.05     433 2748.62     426
 2843.63     433 3041.39     426  3412.2  431.96 3632.22  422.94  3900.8     431
 5491.82  424.94 5550.34  438.94 5690.34  436.94 5754.68     44910010.58     449
10098.15   430.410377.16     41510708.33     41510851.66     43211490.04     426
11769.08     43411796.68     42711808.78     40911852.59  404.6311993.02  433.86
12029.02     42512221.64     43312261.65     44312331.88     44212407.07     447
#Mann= 13 ,-1,0
    1770    .065       0 2623.55     .08       0 2738.05     .05       0
 2843.63    .075       0  3412.2     .04       0  3900.8    .075       0
10010.58    .035       010098.15    .045       010851.66    .085       0
11769.08     .05       011993.02     .09       012221.64     .05       0
12331.88     .08       0
#XS Ineff= 2 , 0
        11769.08     434
Permanent Ineff=
       F       F
Bank Sta=11769.08,11993.02
XS Rating Curve= 0 ,0
Exp/Cntr=0.3,0.1

Type RM Length L Ch R = 1 ,40266   ,72,369,400
XS GIS Cut Line= 3
  2435320.0897576975506.292512432434521.514815036967039.66201472
2434973.482407636962538.86629714
#Sta/Elev= 30
    1833  436.23 2708.07  426.49 2784.41     433 3021.61     432 3093.08     426
  3102.1     433 3416.09     432 3638.88  422.94 3909.11  430.94 5463.09  424.94
 5526.23  439.72 5674.18  437.94 5731.18     449 9986.34     44910069.23   431.8
10171.08  419.2110404.73     41510760.95     42010859.21     43311591.42     425
11760.44     43411794.99     42711814.79     40911848.27  404.6511898.32     410
11970.37  434.6312158.86     42512241.47     44312304.09     44212387.59     447
#Mann= 13 ,-1,0
    1833    .065       0 2784.41     .08       0 3021.61     .05       0
  3102.1    .075       0 3416.09     .04       0 3909.11    .075       0
 9986.34    .035       010069.23    .045       010859.21    .085       0
11760.44     .05       011970.37     .09       012241.47     .05       0
12304.09     .08       0
#XS Ineff= 2 , 0
        11760.44     434
Permanent Ineff=
       F       F
Bank Sta=11760.44,11970.37
XS Rating Curve= 0 ,0
Exp/Cntr=0.3,0.1

Type RM Length L Ch R = 1 ,39914   ,770,362,393
XS GIS Cut Line= 3
  2435324.4372686975505.435307562434528.321817346967040.93154599
2435329.103067376962564.00735618
#Sta/Elev= 30
    1920  434.36 2871.26  432.14  2984.1     426 3002.21     435 3096.04     433
 3380.18  431.96 3659.84  422.94 3900.19     433 5365.38  425.26 5429.85  439.94
  5581.7  437.94 5652.87     449    9901     447 9970.08     43110235.19     417
10634.12     43210926.99     425 11182.7     43311322.61     41711378.85     421
11404.99     43411754.77     433 11808.8  409.7911848.84  404.7111908.49  411.88
11928.47     42911963.39     43312130.81     43312224.97     44212313.56     447
#Mann= 13 ,-1,0
    1920    .065       0 2871.26     .08       0 3002.21     .05       0
 3096.04    .075       0 3380.18     .04       0 3900.19    .075       0
    9901    .035       0 9970.08    .045       010634.12    .085       0
11754.77     .05       011963.39     .09       012130.81     .05       0
12224.97     .08       0
#XS Ineff= 2 , 0
        11754.77     433
Permanent Ineff=
       F       F
Bank Sta=11754.77,11963.39
XS Rating Curve= 0 ,0
Exp/Cntr=0.3,0.1

Type RM Length L Ch R = 1 ,39568   ,22,114,124
XS GIS Cut Line= 3
   2435328.632876975504.561826652434536.119849776967044.36579078
2435673.815162276962615.47400838
#Sta/Elev= 30
    1820  434.95 2502.74  431.35 2688.61  430.72 2871.78     431 3268.76     432
 3554.96  422.94 3750.12  425.94 3776.22     434 5241.23  424.94 5304.13   439.2
  5495.5  438.94 5535.02     449 9770.17     449 9845.39  431.08 9963.51  416.37
10056.41     41610417.15  431.7710842.91     42411053.51     433 11355.1     425
11750.67     434 11779.8     42911802.81     41211858.47  404.7711909.44     411
11929.29     42811975.25     43512022.97     42812083.46     44312221.09   450.5
#Mann= 11 ,-1,0
    1820    .065       0 2502.74     .08       0 2688.61     .05       0
 2871.78    .075       0 3268.76     .04       0 3776.22    .075       0
 9770.17    .035       0 9845.39    .045       010417.15    .085       0
11750.67     .05       011975.25     .08       0
#XS Ineff= 2 , 0
        11750.67     434
Permanent Ineff=
       F       F
Bank Sta=11750.67,11975.25
XS Rating Curve= 0 ,0
Exp/Cntr=0.3,0.1

Type RM Length L Ch R = 1 ,39459   ,251,1297,1406
XS GIS Cut Line= 3
  2435331.6421296975504.218221352434545.059013586967048.95563455
2435784.208319136962635.11014841
#Sta/Elev= 30
    1790  434.85 2478.76  431.54 2675.31     432 2822.41     431 3248.67  430.94
 3520.09  422.94 3715.25  425.94 3738.27     434 5111.95     426 5199.39  431.95
 5203.38  425.65  5263.6  438.94 5459.52  439.22 5498.25     449 9729.32     449
 9809.03     430  9954.7  416.1210312.67  430.6110877.36     42511278.99     432
11349.19     42511389.77     43211752.86     43411787.43  427.1811821.36     408
11861.14  404.79 11918.6     40911938.03     42611986.55  434.1712206.54  452.88
#Mann= 11 ,-1,0
    1790    .065       0 2478.76     .08       0 2675.31     .05       0
 2822.41    .075       0 3248.67     .04       0 3738.27    .075       0
 9729.32    .035       0 9809.03    .045       010312.67    .085       0
11752.86     .05       011986.55     .08       0
#XS Ineff= 2 , 0
         11752.9     434
Permanent Ineff=
       F       F
Bank Sta=11752.86,11986.55
XS Rating Curve= 0 ,0
Exp/Cntr=0.3,0.1

Type RM Length L Ch R = 1 ,38059   ,710,193,200
BEGIN DESCRIPTION:
38059
END DESCRIPTION:
XS GIS Cut Line= 6
2435554.826474776974938.42010256 2435749.6282077  6969102.156369
 2435661.4889483  6965868.123467 2436432.5313695 6965535.1343036
 2436599.6320852 6964389.3009653 2437280.4043457 6962733.3626761
#Sta/Elev= 30
  342.25  438.17  426.76  427.24  615.23  437.76  658.13  429.54 1394.74  430.32
    1444     432  1800.4   431.6    2046  421.65  2288.4   431.6 3533.25  429.56
    3574   438.8    3694   438.8 3734.96  429.15 4277.66     426 4403.05   448.3
    7600     450 7714.85  430.58 7932.69     416 8159.45  417.68 8240.12  428.23
10774.35  433.7110806.32  425.9910823.78     41010862.19     405 10900.6  410.15
10954.14  433.3910955.89     43411148.62     46211221.77   465.311354.83  471.19
#Mann= 12 ,-1,0
  342.25    .065       0 1394.74     .05       0    1444     .08       0
  1800.4     .04       0  2288.4     .08       0    7600    .035       0
 7714.85    .045       0 8240.12      .1       010774.35    .055       0
10954.14    .065       011148.62     .05       011221.77    .065       0
#XS Ineff= 2 , 0
        10774.35  433.71
Permanent Ineff=
       F       F
Bank Sta=10774.35,10955.89
XS Rating Curve= 0 ,0
Exp/Cntr=0.3,0.1

Type RM Length L Ch R = 1 ,37866   ,131,300,300
BEGIN DESCRIPTION:
This cross section corresponds to cross section 37866 of the non-georeferenced CDC model which was the source of this model.
END DESCRIPTION:
XS GIS Cut Line= 6
  2436131.8889326975308.982127732436131.608093226969150.72180648
2436144.560167066969044.508764312436457.089069566966787.15730789
2436742.338827136964727.09154615 2437487.24350536962714.38231698
#Sta/Elev= 30
       0  438.48  1395.6     430 1437.89     421  1560.6     429  1991.1  421.05
  2213.1   425.1 2240.28  431.89 3737.69     428 3772.86     428 3858.86  447.64
    4900  447.64    4900     430 5559.52     428 5589.05     416 5841.23     416
 5899.89  427.69 7189.33     432 7253.33     415  7795.8     415 7864.34   431.2
 7910.54     432 8327.48     426 9005.49     434 9076.68     410  9131.5     405
 9188.45     410 9254.87  434.22 9531.91  459.22 9628.45     463 9710.02  469.46
#Mann= 15 ,-1,0
       0    .065       0  1395.6     .05       0  1560.6     .04       0
 2240.28    .075       0 3737.69    .065       0 3772.86      .1       0
    4900    .085       0 5559.52    .045       0 5899.89    .085       0
 7253.33     .08       0 7910.54    .085       0 9005.49    .055       0
 9254.87    .065       0 9531.91     .05       0 9628.45    .065       0
#XS Ineff= 2 ,-1
       0    7086     434    7086 7876.49   426.5
Permanent Ineff=
       F       T
Bank Sta=9005.49,9254.87
XS Rating Curve= 0 ,0
Exp/Cntr=0.3,0.1

Type RM Length L Ch R = 3 ,37716   ,,,
BEGIN DESCRIPTION:
Hunter Ferrell Road
END DESCRIPTION:
Node Name=Hunter Ferrell R
Bridge Culvert--1,0,-1,-1, 0
Deck Dist Width WeirC Skew NumUp NumDn MinLoCord MaxHiCord MaxSubmerge Is_Ogee
92,115,2.6,0, 17, 17, , , 0.95, 0, 0,0,,
       0     136     336   516.1  1216.1  1316.1  1316.1  1816.1  2316.1  2316.1
  2416.1  2816.1  3116.1  3316.1  3516.1  3716.1  3851.1
   439.5     439     440     439  445.83   446.5   446.5   449.5   446.5   446.5
  445.85  440.68   438.7     440   438.8   440.1  439.29
                                                     440     443     440
       0     136     336  642.15 1342.15 1442.15 1442.15 1942.15 2442.15 2442.15
 2542.15 2942.15 3242.15 3442.15 3642.15 3842.15 3977.15
   439.5     439     440     439  445.83   446.5   446.5   449.5   446.5   446.5
  445.85  440.68   438.7     440   438.8   440.1  439.29
                                                     440     443     440
Pier Skew, UpSta & Num, DnSta & Num=  ,1425.1, 2 ,1529.5, 2 , 0 , 0 , 0 ,,
       3       3
     415     443
       3       3
     415     443
Pier Skew, UpSta & Num, DnSta & Num=  ,1535.1, 2 ,1639.5, 2 , 0 , 0 , 0 ,,
       3       3
     415     443
       3       3
     415     443
Pier Skew, UpSta & Num, DnSta & Num=  ,1607.26, 2 ,1711.66, 2 , 0 , 0 , 0 ,,
       3       3
     415     443
       3       3
     415     443
Pier Skew, UpSta & Num, DnSta & Num=  ,1721.26, 2 ,1825.66, 2 , 0 , 0 , 0 ,,
       3       3
     415     443
       3       3
     415     443
Pier Skew, UpSta & Num, DnSta & Num=  ,1824, 2 ,1928.4, 2 , 0 , 0 , 0 ,,
       3       3
     415     443
       3       3
     415     443
Pier Skew, UpSta & Num, DnSta & Num=  ,1942, 2 ,2046.43, 2 , 0 , 0 , 0 ,,
       3       3
     415     443
       3       3
     415     443
Pier Skew, UpSta & Num, DnSta & Num=  ,2060, 2 ,2164.43, 2 , 0 , 0 , 0 ,,
       3       3
     415     443
       3       3
     415     443
Pier Skew, UpSta & Num, DnSta & Num=  ,2178, 2 ,2282.43, 2 , 0 , 0 , 0 ,,
       3       3
     415     443
       3       3
     415     443
Abutment Skew #Up #Dn= , 2 , 2
  1316.1  1396.1
     440     420
 1442.15 1522.15
     440     420
Abutment Skew #Up #Dn= , 2 , 2
    2236  2316.1
     420     440
 2362.15 2442.15
     420     440
BR Coef=-1 , 0 , 0 ,, 0 ,,,0.8,0,1.2,0,
WSPro=,,,, 1 ,,,, 0 ,,,, 0 ,,,,-1 ,-1 ,-1 , 0 , 0 , 0 , 0 , 0
BC Design=,, 0 ,, 0 ,,,,,,
BC Use User HTab Curves=0
BC User HTab FreeFlow(D)= 0

Type RM Length L Ch R = 1 ,37566   ,172,323,184
BEGIN DESCRIPTION:
---------------------------------------------------------------------
CDC IRV081607-01 Hunter Ferrell Road Improvements
Cross-section 37566 - 41697
---------------------------------------------------------------------
CDC GP083121-1 Hunter-Ferrell Industrial
Located in LOB.
CRoss-sections 37566 - 37866.
Valley storage site.
END DESCRIPTION:
XS GIS Cut Line= 6
  2436329.1844696975557.113521232436354.375036146969200.77288748
2437116.528039386964755.893981982437642.491882476963499.96211064
2437719.336873136963350.069037722438012.404856556962933.11711572
#Sta/Elev= 30
       0  439.26  654.85  430.19  1488.2     432    1547     421    1665     429
  2095.5  420.84  2317.5  424.89 2338.42  430.12 3721.44  428.59 4930.73     430
 5596.53  428.71 5626.32  420.89  5880.7  420.42 5935.55  427.48 5939.87  427.64
 6263.96  429.29    7398     432 7501.49     415 8022.82     415 8102.26  432.17
 9072.14     434 9105.54   428.4 9145.31  409.72 9193.43  405.18 9247.12  410.28
 9309.74  434.14 9591.91  446.82 9746.96   445.8 9822.88  456.88 9842.87  457.38
#Mann= 16 ,-1,0
       0     .07       0  1488.2     .05       0    1665     .04       0
 2338.42    .075       0 3721.44    .065       0 4930.73    .085       0
 5596.53     .05       0 5935.55    .071       0 5939.87    .071       0
 6263.96    .083       0    7398     .08       0 8102.26    .083       0
 9072.14    .055       0 9309.74    .065       0 9746.96     .05       0
 9822.88    .065       0
#XS Ineff= 5 ,-1
       0    3800     434    3800    4948     455    4948 7330.18     434
 7330.18 8102.26   426.5 8102.26 9072.14     434
Permanent Ineff=
       F       F       F       T       F
Bank Sta=9072.14,9309.74
XS Rating Curve= 0 ,0
Exp/Cntr=0.3,0.1

Type RM Length L Ch R = 1 ,37243   ,239,239,239
BEGIN DESCRIPTION:
With fill grading for CDC GP 070319-1.
New cross section
END DESCRIPTION:
XS GIS Cut Line= 6
  2436445.5119926975622.61470257 2436488.91479336969728.51756689
2436740.650838396967575.739720232436740.273542556967255.55302465
2437272.635994886964824.645484892438126.802593636962838.53429964
#Sta/Elev= 30
   -8178   451.7-7646.57  438.05   -4010  431.16   -3998  421.67-3928.02  421.07
-3886.03     431-3223.17  421.95-2972.23  429.96-1506.54  430.35 -694.69  429.49
 -581.71  420.36 -485.73  430.73 -105.83  429.54  595.29  426.46  651.28  416.61
  945.22  416.48  1008.2  429.17 3261.43  427.49 3880.43  436.88 3901.41  434.12
  3943.3  427.84  3975.3  408.25 4028.13  405.36  4093.3  408.41  4173.3  433.77
  4204.3   437.3  4304.3  451.75 4683.37  449.16 4744.83     457 4856.31  463.09
#Mann= 14 ,-1,0
   -8178     .07       0   -4010     .05       0-3886.03     .04       0
-2972.23    .075       0-1506.54    .065       0 -105.83    .085       0
  595.29    .045       0  1008.2    .085       0 3880.43    .055       0
  4204.3    .065       0  4304.3     .09       04551.439    .055       0
 4683.37    .055       0 4744.83    .065       0
#XS Ineff= 4 ,-1
   -8178   -4806     440   -4806 -1593.8  434.12 -1593.8  -242.6     455
  -242.6 3901.41  434.12
Permanent Ineff=
       F       F       F       F
Bank Sta=3901.41,4173.3
XS Rating Curve= 0 ,0
Exp/Cntr=0.3,0.1

Type RM Length L Ch R = 1 ,37015   ,60,160,241
BEGIN DESCRIPTION:
With fill grading for CDC GP 070319-1.
37015
END DESCRIPTION:
XS GIS Cut Line= 6
  2436543.657137 6975906.9500919 2436589.39687586972878.67826131
 2436597.85158336972023.927346142436597.682948476969156.65191273
2437479.554872396964906.894008062438355.561978646962905.79007064
#Sta/Elev= 30
       0  437.84  999.24  430.38 1096.57     426  1690.5     432 1713.73     422
 1743.65     422 1766.01     432 1846.89     434    2800  430.25 4028.45  429.94
 4174.51  423.22    5100  429.33 6241.83     428  6296.2     416  6501.7     416
  6581.7  428.08 8564.02     434 8586.23     440 8882.11     432 9428.39     434
  9459.4     432 9496.32     410    9541   405.5 9587.13     410 9644.33     434
 9714.38  447.26 9769.75  439.02 9847.71  444.9810231.52     44310463.19  460.62
#Mann= 11 ,-1,0
       0     .12       0  999.24     .07       0  1690.5     .05       0
    2800     .12       0    5100    .085       0 6241.83    .045       0
  6581.7     .12       0 9428.39    .055       0 9644.33    .065       0
 9847.71     .09       010231.52     .05       0
#XS Ineff= 4 ,-1
       0     952     440     952    4030     434    4030    5230     455
    5230 9428.39     434
Permanent Ineff=
       F       F       F       F
Bank Sta=9428.39,9644.33
XS Rating Curve= 0 ,0
Exp/Cntr=0.3,0.1

Type RM Length L Ch R = 1 ,36844   ,60,80,94
BEGIN DESCRIPTION:
With fill grading for CDC GP 070319-1.
New cross section
END DESCRIPTION:
XS GIS Cut Line= 6
  2436606.9703316974827.475872892436645.164808886969126.08701323
 2437575.76104486964858.15230764 2438060.13606036963878.98563081
2438192.948458726963782.631492812438570.552690396962988.36077164
#Sta/Elev= 30
   -7020  438.37-4195.64  438.73-3967.75  423.86-3591.93  430.24-3529.96  421.38
-3430.99  433.37 -2820.1   421.9-1678.44  431.66-1573.47  420.28-1552.48  430.08
-1406.52  430.64-1162.91  420.01 -435.88  431.52 -231.08  417.79 -193.11  428.69
  -55.24  430.22  879.36  429.64  1029.3  416.21 1251.21  416.71 1319.18  429.27
 4070.18  433.93 4125.15  430.64 4152.14  409.88 4205.91  405.24 4268.48  408.16
 4303.28  434.98  4322.2  443.56 5044.78     442 5080.76  451.74 5195.73  457.75
#Mann= 11 ,-1,0
   -7020     .12       0-3591.93    .055       0-3430.99     .12       0
33.68994    .085       0970.3198    .045       01305.189    .085       0
 4070.18    .055       04303.279    .065       0  4322.2    .055       0
4438.109     .09       0 5080.76    .065       0
#XS Ineff= 4 ,-1
   -7020 -4280.3     440 -4280.3 -1211.7  433.93 -1211.7   -82.5     455
   -82.5 4070.18  433.93
Permanent Ineff=
       F       F       F       F
Bank Sta=4070.18,4303.28
XS Rating Curve= 0 ,0
Exp/Cntr=0.3,0.1

Type RM Length L Ch R = 1 ,36764   ,165,186,136
BEGIN DESCRIPTION:
With fill grading for CDC GP 070319-1.
New cross section
END DESCRIPTION:
XS GIS Cut Line= 6
  2436663.1047336974830.890236142436699.562994056969060.05663347
2437657.09782438 6964847.04110942438066.820102056963992.87451065
2438299.111632216963761.711259072438628.538794896963013.01328139
#Sta/Elev= 30
   -6955  438.41-4296.36  439.77-3878.43  421.96-3577.48  430.53 -3500.5  421.28
-3432.51   432.9-2763.65  422.02-1682.03  430.83-1608.06  418.86-1298.17   438.3
 -1202.2  419.14-1026.23  438.43 -873.26  423.14 -347.36  430.96 -211.38  418.02
  -148.4  428.97   408.5  429.29  968.19  429.29 1031.17  416.25 1273.12  417.44
 1364.12  429.04 4075.65  434.25 4121.51  408.84 4178.36  405.11 4230.17  408.64
 4265.92  434.48 4280.01  442.77 4308.93  436.99 5067.58  449.03 5186.52  457.04
#Mann= 11 ,-1,0
   -6955     .12       0-3577.48    .055       0-3432.51     .12       0
   408.5    .085       0 1031.17    .045       0 1364.12    .085       0
 4075.65    .055       0 4265.92    .065       0 4280.01    .055       0
 4308.93     .09       0 5067.58    .065       0
#XS Ineff= 4 ,-1
   -6955 -4174.7     440 -4174.7   -1135  434.25   -1135     -50     455
     -50 4075.65  434.25
Permanent Ineff=
       F       F       F       F
Bank Sta=4075.65,4265.92
XS Rating Curve= 0 ,0
Exp/Cntr=0.3,0.1

Type RM Length L Ch R = 1 ,36578   ,75,594,598
BEGIN DESCRIPTION:
With fill grading for CDC GP 070319-1.
New cross section
END DESCRIPTION:
XS GIS Cut Line= 6
  2436704.7713166974825.681913232436736.02125446 6969075.6819303
2437108.383698726967359.37368314 2437920.98673236964770.65215456
2438353.365132636963994.43717156 2438731.83747286963044.78421523
#Sta/Elev= 30
   -6970  439.61-3554.54   430.1-3458.55   421.7-3396.56  433.61-2676.67  421.95
-1672.93  430.76-1585.95  421.01-1535.97  430.95-1497.97   419.1-1265.03  433.82
-1205.05  419.14-1173.07   429.8-1087.11  419.05 -785.26   438.1 -224.53   429.5
 -183.55  416.98 -149.57  428.53  127.29  429.24  1057.9  418.52 1352.85     417
 1404.85  429.79 3951.51  433.52 3964.45  432.73  4022.2  408.18 4082.16  404.82
 4144.67  408.05 4162.59  432.91 4360.45  435.95 5048.93  449.91 5182.83   456.1
#Mann= 10 ,-1,0
   -6970     .12       0-3554.54    .055       0-3396.56     .12       0
  127.29    .085       0  1057.9    .045       0 1404.85    .085       0
 3964.45    .055       0 4162.59    .065       0 4360.45     .09       0
 5048.93    .065       0
#XS Ineff= 4 ,-1
   -6970   -4160     440   -4160   -1146  433.52   -1146-115.669     455
-115.669 3951.51  433.52
Permanent Ineff=
       F       F       F       F
Bank Sta=3951.51,4162.59
XS Rating Curve= 0 ,0
Exp/Cntr=0.3,0.1

Type RM Length L Ch R = 1 ,35984   ,212,407,104
BEGIN DESCRIPTION:
With fill grading for CDC GP 070319-1.
New cross section
END DESCRIPTION:
XS GIS Cut Line= 6
  2436767.2711916974830.890236142436793.312806556969086.09857614
2437167.716913396967332.402280392437996.941632886964851.81537805
2438901.889626136964157.804955072439283.834072226963248.08269314
#Sta/Elev= 30
   -6953  439.04 -3735.6  431.25-3498.61  421.12-3356.61  432.86-2628.63  421.72
-1676.68  430.73-1562.69  419.32-1493.69  430.54-1430.69  420.65 -968.81  430.21
 -847.87  418.43 -806.89  439.94 -738.92   444.5 -550.01  424.96 -232.15  430.51
 -208.16  417.28 -105.21  429.28 1057.32  427.29 1391.27  416.24 1456.27  429.02
 3591.89  428.46 3688.88  428.28  3748.8  406.75 3824.01  403.87 3900.59  407.03
 3932.53  428.87 3975.44  413.75 4013.37  432.02 5148.48  436.28 5350.42  451.88
#Mann= 10 ,-1,0
   -6953     .12       0 -3735.6    .055       0-3356.61     .12       0
-.259765    .085       0 1057.32    .045       0 1456.27    .085       0
 3591.89    .055       0 4013.37    .065       04492.689     .09       0
 5148.48    .065       0
#XS Ineff= 6 ,-1
   -6953 -4088.2     440 -4088.2 -1109.8  428.28 -1109.8  -137.5     455
  -137.5 3688.88  428.28 3932.53  5158.2  428.87  5158.2 5350.42     440
Permanent Ineff=
       F       F       F       F       F       F
Bank Sta=3688.88,3932.53
XS Rating Curve= 0 ,0
Exp/Cntr=0.3,0.1

Type RM Length L Ch R = 1 ,35577   ,111,286,145
BEGIN DESCRIPTION:
With fill grading for CDC GP 070319-1.
New cross section
END DESCRIPTION:
XS GIS Cut Line= 6
  2436855.8130096974825.68191323 2436876.6463013 6969101.7235449
2437239.836847896967560.712191222438231.316492216964988.96831898
2438473.674275226965020.128689722439366.733184646963261.53771873
#Sta/Elev= 30
   -6876  438.44 -3919.3  439.65-3541.37  426.92-3195.43  427.75-1380.06  430.71
-1187.14  421.71 -827.31  430.55 -543.45  417.48 -446.49  432.44 -341.55  417.22
 -293.57  431.16 -155.64  416.69 -104.66  429.54 1154.82  427.64  1194.8  416.75
 1450.76  416.44 1543.76  431.44 3222.59  429.87 3270.57  407.11 3317.84  403.21
 3373.52  406.55 3411.02   431.2 3750.67  440.55 3951.49  437.22 4075.38   417.4
  4355.1  417.56 4390.06   430.8 4537.77  435.96 5160.15     438 5415.94  450.93
#Mann= 10 ,-1,0
   -6876     .12       0-3541.37    .055       0-3195.43     .12       0
1.290039    .085       0 1154.82    .045       0 1543.76    .085       0
 3222.59    .055       0 3411.02     .08       0 4537.77     .09       0
 5160.15     .08       0
#XS Ineff= 6 ,-1
   -6876 -3950.2     440 -3950.2 -1017.1  429.87 -1017.1 -145.48     455
 -145.48 3222.59  429.87 3411.02  5156.9   431.2  5156.95415.939     440
Permanent Ineff=
       F       F       F       F       F       F
Bank Sta=3222.59,3411.02
XS Rating Curve= 0 ,0
Exp/Cntr=0.3,0.1

Type RM Length L Ch R = 1 ,35291   ,119,97,213
BEGIN DESCRIPTION:
With fill grading for CDC GP 070319-1.
New cross section
END DESCRIPTION:
XS GIS Cut Line= 6
   2436951.516236974821.124507652436973.217630486969102.80851647
2438125.992555896965459.743624152438764.013261476964717.55613214
2439202.381479226964088.215855392439497.520324636963293.94513422
#Sta/Elev= 30
   -6793  437.34-3780.83  439.06-3411.87  424.95-2894.91  426.64-2776.92  419.55
-2637.94  426.33 -389.44  431.41 -262.49   430.7  -211.5  416.85 -169.52  427.05
   -2.58  430.16 1235.23  429.48 1291.23  416.46 1531.23  416.56 1589.23  429.68
  2900.3   433.6 2970.29  406.29 3057.21  402.75 3141.25  406.75 3231.23  431.99
 3550.17  439.33 3581.16  437.31 3614.15  418.87 3670.14  416.85 4056.13   417.7
 4181.12  430.81 4259.12  417.69 4362.12  432.21 4498.04  427.51 5345.59  449.35
#Mann= 9 ,-1,0
   -6793     .12       0-2894.91    .055       0-2637.94     .12       0
30.41016    .085       0 1291.23    .045       0 1589.23    .085       0
  2900.3     .05       0 3231.23     .08       04485.061    .075       0
#XS Ineff= 6 ,-1
   -6793 -3804.1     440 -3804.1  -912.7   433.6  -912.7-167.399     455
-167.399  2900.3   433.6 3231.23  4973.2  431.99  4973.2 5345.59     440
Permanent Ineff=
       F       F       F       F       F       F
Bank Sta=2900.3,3231.23
XS Rating Curve= 0 ,0
Exp/Cntr=0.3,0.1

Type RM Length L Ch R = 1 ,35205   ,267,305,178
BEGIN DESCRIPTION:
35205
END DESCRIPTION:
XS GIS Cut Line= 6
  2437023.3251416974807.811870232437086.948046066971651.66234264
2437087.070093056969165.970791732437702.065254146967187.41602181
2438229.261050136965491.521775812439856.698083976963416.27362972
#Sta/Elev= 30
       0     439 1621.39  424.16 1703.39  423.83 3113.89  418.83    3760  426.09
 3940.26     418 3952.48     428  5196.6     428 5244.83     416 5439.96     416
 5518.02     430 6748.51     434 6788.34     408    6857   402.6 6938.95     410
 6984.78     432 7023.02     434 7380.88  437.74 7452.87  416.82  7803.8  418.18
 7845.79  431.45  8114.7   429.6 8169.68   417.9 8276.64  427.58 8297.64  419.73
 8576.54  419.63 8747.49  434.03 9060.37     429 9193.33   450.1 9304.29  446.55
#Mann= 8 ,-1,0
       0     .12       0 1621.39    .055       0 1703.39     .12       0
    3760    .085       0  5196.6    .045       0 5518.02    .085       0
 6748.51    .055       0 7023.02     .08       0
#XS Ineff= 6 ,-1
       0     250     440     250    3706     434    3706    3938     455
    3938 6748.51     434 7334.89    8725     434    8725 9304.29     440
Permanent Ineff=
       F       T       F       F       F       F
#Block Obstruct= 1 ,-1
    3760    3953     428
Bank Sta=6748.51,7023.02
XS Rating Curve= 0 ,0
Exp/Cntr=0.3,0.1

Type RM Length L Ch R = 1 ,34890   ,120,164,157
BEGIN DESCRIPTION:
New cross section
END DESCRIPTION:
XS GIS Cut Line= 6
  2437178.0784416971938.746086062437230.161998476969100.20419098
2437644.658544816967697.86053897 2438612.10346036965468.42438106
2438777.034232816965190.646393312439974.950800236963497.93816456
#Sta/Elev= 30
   -3696  435.54 -3119.7   431.1-2894.78   446.5-2731.84  427.93-2149.03  419.69
-1483.25  432.51-1416.28  422.49-1324.31  439.77-1128.39  422.21  -55.89  416.84
   68.05  429.87 1478.85  429.14 1522.85  418.06 1741.85  416.46 1815.85  431.05
 2870.93  432.67 2909.81  406.64    2957   402.6 3114.18  433.43 3354.46  434.96
 3396.42  417.38 3454.39  430.05 3488.37   417.5 3644.29   418.2 3690.26   431.8
 4876.58   419.4 4998.49  430.93 5221.37  427.27 5367.22  449.48 5434.17  447.36
#Mann= 6 ,-1,0
   -3696     .12       025.07007    .085       0 1478.85    .045       0
 1815.85    .085       0 2870.93    .055       0 3114.18     .08       0
#XS Ineff= 6 ,-1
   -3696 -3454.7     440 -3454.7-649.399  432.67-649.399    -219     455
    -219 2870.93  432.67 3114.18  4796.7  433.43  4796.7 5434.17     440
Permanent Ineff=
       F       F       F       F       F       F
Bank Sta=2870.93,3114.18
XS Rating Curve= 0 ,0
Exp/Cntr=0.3,0.1

Type RM Length L Ch R = 1 ,34726   ,23,468,565
BEGIN DESCRIPTION:
New cross section
END DESCRIPTION:
XS GIS Cut Line= 6
  2437347.3494286971951.766729312437373.391042726969152.28774823
2437685.989498886967883.628868222438586.061845726965824.32721256
2439402.034295146964687.174303142440079.117586646963550.02139373
#Sta/Elev= 30
   -3615  436.31-3145.47  430.16-2766.52  443.47-2762.52   429.6-1999.63  419.37
-1515.69  436.65-1384.71  422.36 -229.99  419.81  -99.04  431.44  -40.06   418.6
  139.88   429.3  214.86  416.66  274.83  428.44 1581.49  426.21 1828.42  416.16
  1910.4   430.8 2826.16  432.68 2873.15   406.5    2927   402.6 2997.14  406.97
 3056.14  433.73 3139.93  420.21 3323.91  432.78  3430.9  416.94 3571.89   418.6
 3612.89  430.64 5014.43  419.48  5080.6  430.14 5266.43  426.56 5463.41  447.78
#Mann= 6 ,-1,0
   -3615     .12       030.91992    .085       0 1581.49    .045       0
  1910.4    .085       0 2826.16    .055       0 3056.14     .08       0
#XS Ineff= 6 ,-1
   -3615 -3260.6     440 -3260.6    -530  432.68    -530  -136.6     455
  -136.6 2826.16  432.68 3056.14  4775.9  433.73  4775.9 5463.41     440
Permanent Ineff=
       F       F       F       F       F       F
Bank Sta=2826.16,3056.14
XS Rating Curve= 0 ,0
Exp/Cntr=0.3,0.1

Type RM Length L Ch R = 1 ,34268   ,660,886,300
BEGIN DESCRIPTION:
STATIONS 7543-7573 ADDED FROM EFFECTIVE SECTION
FOR FLOWLINE
END DESCRIPTION:
XS GIS Cut Line= 6
  2437489.2313626971974.344768152437489.392779226969177.58034857
 2437700.49504736968636.177888072438650.537110466966217.65286948
2439213.273845886965876.417987642440272.360966556963674.98177373
#Sta/Elev= 30
    1249     440 1632.15  434.35 2101.28     440 2242.11  429.14 2793.01     422
 4627.69  423.24 5155.75     418 5197.43     428 5269.62     418 5325.11     428
 6507.97     430    6571     416 6769.38     416 6844.63     432 7393.73     432
 7470.61     430 7506.88     408    7543   402.6 7636.07  431.81 7639.87     434
 7730.86   435.3 7781.41   423.2 7981.54  434.53 8071.49  420.02 8366.35  430.89
 8593.24  422.31 9732.67  419.4310281.94 430.03510288.54  441.0810333.35     442
#Mann= 8 ,-1,0
    1249     .12       0 1632.15      .1       0 4627.69      .1       0
 6507.97    .045       0 6844.63      .1       0 7393.73    .055       0
 7639.87    .075       010281.94     .05       0
#XS Ineff= 6 ,-1
    1249 2101.28     440 2101.28    4389     430 4389.04 4626.26     445
 4626.26    6844     430    7639    9600     430    960010326.63 440.463
Permanent Ineff=
       F       F       T       F       F       F
Bank Sta=7393.73,7636.07
XS Rating Curve= 0 ,0
Exp/Cntr=0.3,0.1

Type RM Length L Ch R = 1 ,33382   ,56,47,10
BEGIN DESCRIPTION:
33382
END DESCRIPTION:
XS GIS Cut Line= 6
  2438291.2596136971935.470830142438326.285462386970426.81308632
2438292.569322476969094.10052864 2438626.77075386967522.91994397
2439270.00011039 6966664.41313082440310.726375396963618.04455164
#Sta/Elev= 30
    4895  439.03 5626.66  427.69  5799.9     439 6199.87  433.68 6253.14  422.11
 6654.71  422.63 8482.86     416 8628.25  417.03  8687.4  429.99 8732.44     416
 8775.09     42810039.77  430.8810091.57     406   10160   402.510229.52  407.87
10283.96     43211016.26  431.2711055.24  423.7811326.15  432.6811427.12  420.18
11558.08   420.111592.06  429.7811696.03   430.811861.92  422.1113125.92  420.77
13580.27430.456313585.75  430.8413589.74     44213647.01  448.2113676.11   447.6
#Mann= 8 ,-1,0
    4895    .085       0  5799.9      .1       0 6199.87    .085       0
 6654.71     .12       010039.77    .055       010283.96    .075       0
13580.27     .05       013647.01    .075       0
#XS Ineff= 4 ,-1
    4895 5874.95     440    6137    9895     430   1028312823.14     430
12823.14   13636     440
Permanent Ineff=
       T       F       F       F
Bank Sta=10039.77,10283.96
XS Rating Curve= 0 ,0
Exp/Cntr=0.3,0.1

Type RM Length L Ch R = 1 ,33335   ,55,22,13
BEGIN DESCRIPTION:
33335
END DESCRIPTION:
XS GIS Cut Line= 6
  2438405.4798576971935.231329312438437.076579396970272.24712248
 2438395.84405036969130.753998642438688.812624476967524.85104248
2439284.515829386966668.731363642440320.431736566963618.92676772
#Sta/Elev= 30
       0  440.75  685.59  434.78  721.21  427.12  764.15  438.94  987.68  439.45
 1297.84     440 1346.95  426.21 1373.92  430.01    1653     423 3354.07     418
 3751.43  416.84 3771.72     428 3803.44     416  3832.1   416.7 3840.67     428
 5068.05  431.67 5115.05     406    5188   402.3 5261.81   407.7 5291.99     428
 5337.17     432 6104.16   425.5 6355.08  433.18 6496.06  420.19 6737.02  430.64
 6802.01  422.77 8206.53  420.09 8596.03  428.27 8683.95  446.05 8727.41  447.35
#Mann= 9 ,-1,0
       0    .085       0  987.68      .1       0 1373.92    .085       0
    1653    .085       0 3354.07     .12       0 5068.05    .055       0
 5337.17    .075       0 8596.03     .05       0 8683.95    .075       0
#XS Ineff= 4 ,-1
       0 1042.63     440    1288    4867     430    5337    7857     430
    7857    8667     440
Permanent Ineff=
       T       F       F       F
Bank Sta=5068.05,5337.17
XS Rating Curve= 0 ,0
Exp/Cntr=0.3,0.1

Type RM Length L Ch R = 1 ,33313   ,50,19,13
BEGIN DESCRIPTION:
33313
STATIONS 1060-1532 2009 CGP TOPOGRAPHY
END DESCRIPTION:
XS GIS Cut Line= 6
  2438449.0834456971937.828765062438492.486245476970352.54223748
2438502.251973976969218.644570892438747.477533396967524.85104248
2439295.437723556966671.986606482440324.843145066963618.92676772
#Sta/Elev= 30
       0  442.66  650.49  431.47 1007.64  439.76    1326     433    1370     422
 1852.02     424 3390.11     418 3742.22  416.99  3754.7     428 3788.34     416
 3852.63     428 4163.98  416.06 4230.62     428 5029.25  431.35 5071.39     406
    5144   402.2  5217.9   407.3 5256.99     428 5302.07     432 6020.97  432.68
 6103.89  424.65 6313.68  433.14 6508.54  420.04 6561.51  429.55 6691.44  430.21
 6765.41  422.91 8170.51  420.44 8554.25  428.12 8645.86  446.65 8689.03  447.31
#Mann= 9 ,-1,0
       0    .085       0 1007.64      .1       0    1326    .085       0
 1852.02    .085       0 3390.11     .12       0 5029.25    .055       0
 5302.07    .075       0 8554.25     .05       0 8645.86    .075       0
#XS Ineff= 4 ,-1
       0 1040.76     440    1325    4795     430    5795 7812.07     430
 7812.07    8627     440
Permanent Ineff=
       T       F       F       F
#Block Obstruct= 1 ,-1
    3770    3839     426
Bank Sta=5029.25,5302.07
XS Rating Curve= 0 ,0
Exp/Cntr=0.3,0.1

Type RM Length L Ch R = 1 ,33294   ,42,27,25
BEGIN DESCRIPTION:
33294
STATIONS 1041-1614 2009 CGP TOPOGRAPHY
END DESCRIPTION:
XS GIS Cut Line= 6
  2438466.3977146971932.283172472438536.901182896969172.12694739
2438759.470619636967536.536714642439148.939656976966922.79351956
2439316.339584636966666.023363812440325.204364816963620.20858932
#Sta/Elev= 30
       0  442.98  647.85  431.58  987.02  439.76 1304.11     439    1368     422
    2008     420  3310.3  416.73 3732.68  416.43 3759.42     430 3786.24     416
 3874.24   424.6  3967.7  416.06 4017.49  425.41  4120.3     416 4216.51     428
 4996.94   431.7 5030.93     406  5098.5   402.1 5167.67  406.06 5217.83     428
  5266.5     432 5982.48   431.2  6067.4  423.05 6262.85  433.24 6457.91  420.07
 6527.91  429.99  8151.9   420.5  8519.5  428.11 8608.24  445.98 8651.96  447.33
#Mann= 9 ,-1,0
       0    .085       0  987.02      .1       0    1368    .085       0
    2008    .085       0  3310.3     .12       0 4996.94    .055       0
  5266.5    .075       0  8519.5     .05       0 8608.24    .075       0
#XS Ineff= 4 ,-1
       0 1008.91     440    1322    4814     430    5795 7771.64     430
 7771.64 8651.96     440
Permanent Ineff=
       T       F       F       F
#Block Obstruct= 1 ,-1
    3398    4017     422
Bank Sta=4996.94,5266.5
XS Rating Curve= 0 ,0
Exp/Cntr=0.3,0.1

Type RM Length L Ch R = 1 ,33267   ,42,47,25
BEGIN DESCRIPTION:
33267
STATIONS 1027-1778 2009 CGP TOPOGRAPHY
END DESCRIPTION:
XS GIS Cut Line= 6
  2438482.6266856971933.408498322438526.897593986970412.57525389
2438571.168174716969087.054282892438774.293424646967542.78342131
2439328.980635466966672.991853822440325.725689226963620.69152798
#Sta/Elev= 30
       0  443.06  633.43  433.53  932.94  439.17 1294.16     439    1365     422
    1505     423    1636     423 3311.17  417.72 3732.06  416.49    3756     430
 3804.84     416  3921.5   416.3 3954.56     426 4085.74     416  4204.4     428
 4990.42  431.55 5019.67     406    5080   402.1 5255.59     432 5974.91  431.67
 6008.66  423.31 6259.84  433.17 6434.59  422.72 6521.96  429.92 6820.79  422.23
    8478  427.54 8538.01  428.93 8554.67  442.03 8602.72  446.25 8645.26  447.34
#Mann= 10 ,-1,0
       0    .085       0  932.94      .1       0    1365    .085       0
    1505    .085       0    1636    .085       0 3311.17     .12       0
 4990.42    .055       0 5255.59    .075       0    8478     .05       0
 8602.72    .075       0
#XS Ineff= 4 ,-1
       0  997.87     440    1301    4782     430    5645 7760.12     430
 7760.12    8580     440
Permanent Ineff=
       T       F       F       F
#Block Obstruct= 1 ,-1
    3378    3953     424
Bank Sta=4990.42,5255.59
XS Rating Curve= 0 ,0
Exp/Cntr=0.3,0.1

Type RM Length L Ch R = 1 ,33220   ,63,32,20
BEGIN DESCRIPTION:
33220
STATIONS 1018-1847 2009 CGP TOPOGRAPHY
END DESCRIPTION:
XS GIS Cut Line= 6
   2438532.237156971926.218223972438601.681565146969031.25321339
2438801.33438106 6967542.53768692439387.271857476966661.46136506
2440174.614442886964094.320830062440326.789663466963622.57078931
#Sta/Elev= 30
       0  441.98  647.03   430.4  959.21  439.59 1289.39     439    1362     422
    1508     423    1639     421    2180     420 3297.73  417.62 3390.82  423.64
 3412.93     414 3508.32  414.49 3554.53     426 3720.65  417.58 3767.38  428.66
 4067.54  416.19 4089.48     426 4179.87     428 4988.64  431.81 5016.95     406
    5073   401.9 5242.89     432 5964.24  431.45 6028.89  422.93 6272.57  433.23
 6805.69  422.36 8506.55   428.1 8543.01  430.89 8548.95  442.04 8635.78  447.42
#Mann= 11 ,-1,0
       0    .085       0  959.21      .1       0    1362    .085       0
    1508    .085       0    1639    .085       0    2180    .085       0
 3297.73     .12       0 4988.64    .055       0 5242.89    .075       0
 8506.55     .05       0 8635.78    .075       0
#XS Ineff= 4 ,-1
       0  997.95     440    1320    4853     430    5243 7744.36     430
 7744.36 8635.78     440
Permanent Ineff=
       T       F       F       F
#Block Obstruct= 1 ,-1
    3362    3737     424
Bank Sta=4988.64,5242.89
XS Rating Curve= 0 ,0
Exp/Cntr=0.3,0.1

Type RM Length L Ch R = 1 ,33188   ,118,52,25
BEGIN DESCRIPTION:
33188
STATIONS 1015-1794, 2009 CGP TOPOGRAPHY
END DESCRIPTION:
XS GIS Cut Line= 6
  2438555.1209626971901.796684892438606.02177955 6970289.9337669
2438627.723179716969083.336442562438857.75815272 6967542.5376869
2439413.313472056966670.142121972440331.151531386963676.44371305
#Sta/Elev= 30
       0  441.78  647.84  430.66  726.52  439.08  985.59   439.9 1292.69     439
    1359     422    2205     420  3271.2  416.05 3321.97  416.01 3352.08     426
 3414.85     414 3516.09  425.95    3572     414 3639.22     426 3833.73  425.68
 3880.52     416 4030.41  427.81 4973.02  430.79 5009.14     406    5061   401.7
 5230.03     432 5952.02  430.33 5999.99  422.62 6231.86  433.25 6872.06  422.38
 8359.79   422.4 8503.88  429.25 8513.87  431.74 8516.87  442.75 8553.83  443.81
#Mann= 7 ,-1,0
       0    .085       0  985.59      .1       0    1359    .085       0
    2205    .085       0  3271.2     .12       0 4973.02    .055       0
 5230.03    .075       0
#XS Ineff= 4 ,-1
       0  998.33     440    1320    4973     430    5230 7689.76     430
 7689.76 8553.79     440
Permanent Ineff=
       T       F       F       F
#Block Obstruct= 1 ,-1
    3352    3639     426
Bank Sta=4973.02,5230.03
XS Rating Curve= 0 ,0
Exp/Cntr=0.3,0.1

Type RM Length L Ch R = 1 ,33136   ,184,74,25
BEGIN DESCRIPTION:
33136 The reach length has been updated and it is the same with the 2018 georeferenced model.
STATIONS 1024-1873 2009 CGP TOPOGRAPHY
END DESCRIPTION:
XS GIS Cut Line= 6
2438590.401075886972015.513649062438673.477025236969220.41687706
2438763.768183226968538.219094492438941.706147556967577.18755198
2439436.497808896966676.146046982440386.298074636963652.28693722
#Sta/Elev= 30
       0  440.86  649.96  431.08  722.97   439.4   921.6     439 1295.79     439
    1352     422 2261.87  420.29 3241.53  416.28 3327.43     426 3393.52  424.76
 3421.65     414 3460.22     426 3586.96  425.95 3674.75     414  3729.4  423.52
 3752.83     414  3869.9  426.75 4957.16  431.07 4997.22     406    5048   401.6
 5226.59     432 5924.98  428.69  5945.4     420 6190.62     434  6617.3  429.62
 6646.77     422  8423.1  427.31  8483.3     442  8530.5  442.74 8559.47     448
#Mann= 9 ,-1,0
       0    .085       0   921.6      .1       0    1352    .085       0
 2261.87    .085       0 3241.53     .12       0 4957.16    .055       0
 5226.59    .075       0  8423.1     .05       0  8530.5    .075       0
#XS Ineff= 4 ,-1
       0  996.56     440    1300    4815     430    5227    7618     430
    7618    8520     440
Permanent Ineff=
       T       F       F       F
#Block Obstruct= 1 ,-1
    3327    3717   423.6
Bank Sta=4957.16,5226.59
XS Rating Curve= 0 ,0
Exp/Cntr=0.3,0.1

Type RM Length L Ch R = 1 ,33062   ,190,48,20
BEGIN DESCRIPTION:
33062 The reach length has been updated and it is the same with the 2018 georeferenced model.
STATIONS 1073-1948 2009 CGP TOPOGRAPHY
END DESCRIPTION:
XS GIS Cut Line= 6
2438646.363562396971916.28386064 2438699.51863986970095.41676748
2438748.997871556969314.167017642439051.081256886967600.62516914
2439478.164392226966699.583664152440365.240632846963740.73208122
#Sta/Elev= 30
       0  440.32  693.06  432.63  918.36     439 1292.59  438.98    1350     422
    1531     422 1747.74   422.2 2458.68   418.5 3215.26  416.83 3269.16     426
 3391.74  424.83 3426.82     414 3538.61  425.96 3571.63     414  3608.2  414.51
 3623.64  426.08 4620.26  429.87 4718.72  418.82 4816.56  431.82 4929.56  431.48
 4958.48     406    5002   401.3 5096.21     408 5187.05     432 5885.88  428.62
 5907.44     420 6173.44  433.48 6606.15     422 8378.48  427.15 8431.47     440
#Mann= 12 ,-1,0
       0    .085       0  918.36      .1       0    1350    .085       0
    1531    .085       0 1747.74    .085       0 2458.68    .085       0
 3215.26     .12       0 4620.26    .055       0 4816.56     .07       0
 4929.56    .055       0 5187.05    .075       0 8378.48     .05       0
#XS Ineff= 5 ,-1
       0  993.31     440    1300    4600     430    4600    4900     430
    5187    7559     430    7559 8431.47     440
Permanent Ineff=
       T       F       T       F       F
#Block Obstruct= 1 ,-1
    3269 3533.41     426
Bank Sta=4929.56,5187.05
XS Rating Curve= 0 ,0
Exp/Cntr=0.3,0.1

Type RM Length L Ch R = 1 ,33014   ,60,47,24
BEGIN DESCRIPTION:
33014 The reach length has been updated and it is the same with the 2018 georeferenced mode.
STATIONS 1059-1985 2009 CGP TOPOGRAPHY
END DESCRIPTION:
XS GIS Cut Line= 6
2438846.289343646972015.82434398 2438845.87267786969631.35437539
2438997.695536886968443.333457482439178.685332396967561.56258322
2439501.602009396966702.187661562440395.831192056963661.45358557
#Sta/Elev= 30
       0  438.85  910.52     439 1284.78     439    1343     422    1515     423
    1767     421    2022   418.7 3092.42  416.45 3203.19     426 3408.66     424
 3461.08     414 3546.68  414.65 3579.51     426 4369.25  429.97  4558.4     412
 4684.81     412 4769.52  431.75 4884.41  431.44 4919.89     406    4966   401.1
 5070.81     408 5136.79     432 5836.33  429.29 5893.81  419.08 5939.06  429.67
 6127.95  432.55  6554.5     422 8328.81  427.08 8442.69     443 8471.68     448
#Mann= 13 ,-1,0
       0    .085       0  910.52      .1       0    1343    .085       0
    1515    .085       0    1767    .065       0    2022    .085       0
 3092.42     .12       0 4369.25    .055       0 4769.52     .07       0
 4884.41    .055       0 5136.79    .075       0 8328.81     .05       0
 8442.69    .075       0
#XS Ineff= 5 ,-1
       0  985.48     440    1300    4350     430    4350    4780     430
    5137    7516     430    7516    8432     440
Permanent Ineff=
       T       F       T       F       F
Bank Sta=4884.41,5136.79
XS Rating Curve= 0 ,0
Exp/Cntr=0.3,0.1

Type RM Length L Ch R = 1 ,32967   ,54,48,60
BEGIN DESCRIPTION:
32967 The reach length has been updated and it is the same with the 2018 georeferenced model.
STATIONS 6649-7540 2009 CGP TOPOGRAPHY
END DESCRIPTION:
XS GIS Cut Line= 6
2438854.218789736972396.935130312438900.039564226970957.39601465
2438905.247887136969452.187738982439173.477009486967777.70847639
2439514.622980716966785.521156312440441.649341886963559.06993206
#Sta/Elev= 30
    5308  438.92 6234.57     439 6578.74     440    6643     423    6943     421
    7109     420    7372   418.7 8365.91  416.14  8655.9  414.02    8846  425.97
 8903.09     414  9010.2  414.73 9024.68     426 9082.24     428 9484.89  430.12
 9712.35     412 9989.64     412   10071   431.610175.69  431.2710210.15     406
   10273     40110377.47     40810428.55     43211135.59  429.48 11159.4     418
11309.65     43211840.67     42213625.75  427.1513737.19     44313897.58  443.68
#Mann= 13 ,-1,0
    5308    .085       0 6234.57      .1       0    6643    .085       0
    6943    .085       0    7109    .065       0    7372    .085       0
 8365.91     .12       0 9484.89    .055       0   10071     .07       0
10175.69    .055       010428.55    .075       013625.75     .05       0
13737.19    .075       0
#XS Ineff= 5 ,-1
    5308 6309.43     440    6610    9480     430    9480   10100     430
   10683   12779     430   12779   13731     440
Permanent Ineff=
       T       F       T       F       F
#Block Obstruct= 1 ,-1
    8512    8689     426
Bank Sta=10175.69,10428.55
XS Rating Curve= 0 ,0
Exp/Cntr=0.3,0.1
